HEC-RAS study ozz_def.prj: ozzeri

--- ozz_def.g04 (geometry) --- (continued)

Type RM Length L Ch R = 1 ,782     ,123.031,123.031,123.031
XS GIS Cut Line= 3
      5315453.94      15922360.7      5315572.64     15922571.92
      5315572.64     15922571.92
#Sta/Elev= 19
       0  44.455   2.395  44.921    2.48  46.578  15.335  45.381  26.693  38.228
  39.701  36.348  44.692  31.837  50.577   31.07  62.106  30.896  66.135  30.869
  73.002   31.02  80.036  30.709  89.961  30.571  96.982  31.588 103.458  35.692
  113.75  35.879 127.024   44.36 144.249  44.436 242.756  41.703
#Mann= 3 , 0 , 0
       0    .035       0   2.395    .035       0 144.249    .035       0
Bank Sta=2.395,144.249
XS Rating Curve= 0
Exp/Cntr=.3,.1

Type RM Length L Ch R = 1 ,781     ,77.493,77.493,77.493
XS GIS Cut Line= 2
      5315354.92      15922412.2      5315421.33     15922556.76
#Sta/Elev= 15
       0  46.158  10.781  45.197  22.008  38.041   34.79  36.368  39.419  32.142
  47.283   31.03  55.774  31.142  65.804    30.2  75.591  30.531  82.749  30.049
  87.385  30.394  93.297  31.214 110.328  32.769 143.058  34.321 162.129  34.961
#Mann= 3 , 0 , 0
       0    .035       0       0    .035       0 162.129    .035       0
Bank Sta=0,162.129
XS Rating Curve= 0
Exp/Cntr=.3,.1

Type RM Length L Ch R = 1 ,780     ,29.528,29.528,29.528
XS GIS Cut Line= 2
      5315283.07     15922441.17      5315322.51     15922548.92
#Sta/Elev= 16
       0  44.911   7.799   44.61  20.512  36.365  29.429  35.361  35.689  32.037
  42.037  32.402   48.55  32.395  54.377  32.392  62.828  32.402  71.772  32.408
   82.48  32.431  88.051  32.451  92.264  31.211  94.167  34.541 105.725  38.071
 115.577  43.143
#Mann= 3 , 0 , 0
       0    .035       0       0    .035       0 115.577    .035       0
Bank Sta=0,115.577
XS Rating Curve= 0
Exp/Cntr=.3,.1

Type RM Length L Ch R = 3 ,779.5   ,,,
BEGIN DESCRIPTION:
Ponte di Pontetetto
END DESCRIPTION:
Bridge Culvert--1,0,-1,-1, 0
Deck Dist Width WeirC Skew NumUp NumDn MinLoCord MaxHiCord MaxSubmerge Is_Ogee
1.64,26.247,2.61,0, 19, 19, , , .95, 0, 0,0,,
       0   7.776  20.472  24.934  29.396  35.663  40.092  42.159   51.64  54.331
  62.762  71.686  73.097  82.349  87.238   91.47   93.34 105.741 115.584
  45.932  45.932  45.932  45.932  45.932  45.932  45.932  45.932  45.932  45.932
  45.932  45.932  45.932  45.932  45.932  45.932  45.932  45.932  45.932
  44.915  44.619  36.352  41.831  42.913  41.634  40.387  31.234  30.741  40.354
   42.52  38.353  30.741  30.512  40.945  42.421  42.651  38.058  43.143
       0   7.776  20.472  24.934  29.396  35.663  40.092  42.159   51.64  54.331
  62.762  71.686  73.097  82.349  87.238   91.47   93.34 105.741 115.584
  45.932  45.932  45.932  45.932  45.932  45.932  45.932  45.932  45.932  45.932
  45.932  45.932  45.932  45.932  45.932  45.932  45.932  45.932  45.932
  44.915  44.619  36.352  41.831  42.913  41.634  40.387  31.234  30.741  40.354
   42.52  38.353  30.741  30.512  40.945  42.421  42.651  38.058  43.143
BR Coef=-1 , 0 , 0 ,1.25, 0 ,,,.8,-1,2,0,
WSPro=,,,, 1 ,,,, 0 ,,,, 0 ,,,,-1 ,-1 ,-1 , 0 , 0 , 0 , 0 , 0
BC Design=,, 0 ,, 0 ,,,,,,
BC HTab Sub Flow Pts= 40

Type RM Length L Ch R = 1 ,779.3   ,29.856,29.856,29.856
XS GIS Cut Line= 2
      5315283.07     15922441.17      5315322.51     15922548.92
#Sta/Elev= 16
       0  44.911   7.799   44.61  20.512  36.365  29.429  35.361  35.689  32.037
  42.037  32.402   48.55  32.395  54.377  32.392  62.828  32.402  71.772  32.408
   82.48  32.431  88.051  32.451  92.264  31.211  94.167  34.541 105.725  38.071
 115.577  43.143
#Mann= 3 , 0 , 0
       0    .035       0       0    .035       0 115.577    .035       0
Bank Sta=0,115.577
XS Rating Curve= 0
Exp/Cntr=.3,.1

Type RM Length L Ch R = 1 ,779     ,62.566,62.566,62.566
XS GIS Cut Line= 3
      5315249.61      15922433.1      5315296.72     15922565.12
      5315296.72     15922565.12
#Sta/Elev= 14
       0  37.756   18.72  43.445  18.819  46.427  20.118  46.444  20.899  32.789
  37.572  33.114  68.642  31.686  77.703  30.423   88.74  31.385 102.159  31.043
 107.874  31.394  111.66  34.636 128.816  37.359 140.656  44.442
#Mann= 3 , 0 , 0
       0    .035       0       0    .035       0 140.656    .035       0
Bank Sta=0,140.656
XS Rating Curve= 0
Exp/Cntr=.3,.1

Type RM Length L Ch R = 6 ,778.55  ,,,
Lateral Weir Pos= 0
Lateral Weir End=                ,                ,        ,c14
Lateral Weir Distance=3.281
Lateral Weir WD=9.843
Lateral Weir Coef=3.01
Lateral Weir Is Ogee= 0
Lateral Weir WSCriteria=-1
Lateral Weir SE= 6
       0   49.21    3.28   49.21    3.28   43.61  167.32   43.61  167.32   49.21
   170.6   49.21

Type RM Length L Ch R = 1 ,778.5   ,123.392,123.392,123.392
XS GIS Cut Line= 2
      5315198.98     15922469.23      5315235.14     15922594.82
#Sta/Elev= 21
       0  46.749     .23  43.182  15.226  42.897  20.659  37.884  33.396   37.07
  38.845   34.37  41.493  32.201  46.588  29.875  57.618    29.4  72.503  29.511
  81.936  29.213  89.688  30.814  91.486  32.169 100.148  36.827 110.075  37.014
 120.036  43.107 123.189  43.885 129.665  44.665  130.03  45.443 130.807  45.479
 131.201  42.543
#Mann= 3 , 0 , 0
       0    .035       0       0    .035       0 131.201    .035       0
Bank Sta=0,131.201
XS Rating Curve= 0
Exp/Cntr=.3,.1

Type RM Length L Ch R = 1 ,778     ,149.18,149.18,149.18
XS GIS Cut Line= 2
      5315073.69     15922487.24      5315175.89     15922785.96
#Sta/Elev= 19
       0   43.75  26.972   43.78  39.252  43.576  46.345  37.818  56.972  37.421
  63.255  34.459  64.754  31.877  71.739  31.772  81.283  31.296  89.383  31.627
   99.14  31.296 109.452  30.988 115.997  30.784  119.16   33.97 129.465   38.72
 146.214  44.072 154.213  44.662 162.198  42.772 315.945  41.795
#Mann= 3 , 0 , 0
       0    .035       0       0    .035       0 315.945    .035       0
Bank Sta=0,315.945
XS Rating Curve= 0
Exp/Cntr=.3,.1

Type RM Length L Ch R = 1 ,777     ,172.736,172.736,172.736
XS GIS Cut Line= 2
       5314931.4     15922518.31      5315014.07     15922788.75
#Sta/Elev= 18
       0  44.022  54.639   43.74  63.317  38.123   76.24  37.116  83.642  32.297
  89.117  30.961  98.993  31.932 106.355  31.627  119.37  31.598 127.119  30.909
 134.442  30.561 136.965   32.89 146.358  38.596 155.758  39.147 163.445  43.684
 171.565   44.57  174.76  42.398 283.465  41.342
#Mann= 3 , 0 , 0
       0    .035       0       0    .035       0 283.465    .035       0
Bank Sta=0,283.465
XS Rating Curve= 0
Exp/Cntr=.3,.1

Type RM Length L Ch R = 1 ,776     ,347.966,347.966,347.966
XS GIS Cut Line= 2
      5314764.24     15922596.03      5314784.71     15922646.82
#Sta/Elev= 18
       0  44.905  15.689  45.531  35.108  45.249  44.938  38.963  57.884  37.772
  66.677  32.297   75.19  31.808  82.152  31.808  95.197  31.814 108.579  31.257
  116.65  30.856 118.839  33.245 128.619  37.989 139.951  38.921 148.084  43.297
 153.504  43.904 158.917  40.548 262.992  40.748
#Mann= 3 , 0 , 0
       0    .035       0       0    .035       0 262.992    .035       0
Bank Sta=0,262.992
XS Rating Curve= 0
Exp/Cntr=.3,.1

Type RM Length L Ch R = 1 ,775     ,243.898,243.898,243.898
XS GIS Cut Line= 3
      5314438.16     15922721.19      5314683.89      15922793.8
      5314683.89      15922793.8
#Sta/Elev= 20
       0    45.2  16.778  44.925  20.994  44.108  30.633  43.727  38.704  38.789
   51.67  37.467  60.807  32.405  61.434   31.47  69.075  30.781  82.976   30.65
  94.186  30.223 104.547  30.259 111.325  30.075 114.957  32.963 125.843  38.251
 134.229  38.491 143.353  42.828 148.878  42.972 155.925  40.915 184.682  40.653
#Mann= 3 , 0 , 0
       0    .035       0       0    .035       0 143.353    .035       0
Bank Sta=0,143.353
XS Rating Curve= 0
Exp/Cntr=.3,.1

Type RM Length L Ch R = 6 ,773.555 ,,,
Lateral Weir Pos= 0
Lateral Weir End=                ,                ,        ,c12
Lateral Weir Distance=3.281
Lateral Weir WD=9.843
Lateral Weir Coef=3.01
Lateral Weir Is Ogee= 0
Lateral Weir WSCriteria=-1
Lateral Weir SE= 6
       0   49.21    3.28   49.21    3.28   43.61      36   43.61      36   49.21
      40   49.21

Type RM Length L Ch R = 6 ,773.55  ,,,
Lateral Weir Pos= 3
Lateral Weir End=                ,                ,        ,c11
Lateral Weir Distance=3.281
Lateral Weir WD=9.843
Lateral Weir Coef=3.01
Lateral Weir Is Ogee= 0
Lateral Weir WSCriteria=-1
Lateral Weir SE= 6
       0   49.21    3.28   49.21    3.28   42.62  331.37   42.62  331.37   49.21
  334.65   49.21

Type RM Length L Ch R = 1 ,773     ,224.705,224.705,224.705
XS GIS Cut Line= 3
      5314213.12     15922725.43      5314269.85     15922983.07
      5314269.85     15922983.07
#Sta/Elev= 18
       0  43.543  59.633  43.976  65.797  42.579  77.008  37.543  90.525  35.679
  96.588  33.031  97.313  31.969 105.348  31.532 115.344  31.322  126.22  31.339
 137.946  30.545 148.583  31.001 156.975  31.457 161.355  35.968 172.621  37.178
 182.651  43.159 210.443  42.648 263.858  42.254
#Mann= 3 , 0 , 0
       0    .035       0       0    .035       0 263.858    .035       0
Bank Sta=0,263.858
XS Rating Curve= 0
Exp/Cntr=.3,.1

Type RM Length L Ch R = 1 ,772.5   ,40.354,40.354,40.354
#Sta/Elev= 27
       0  53.169   20.83  54.803  38.891  54.482  46.955  48.625  53.888  43.097
  59.383  42.644  68.583  37.113  81.821  36.522  88.671  33.219  90.577  32.051
  92.539  31.037  98.255  30.827 101.516  29.052 110.325  27.871 119.879  27.549
 129.662  27.477 137.917   27.27 145.144  30.676 146.631   31.27 147.776  32.037
 153.333  36.266 153.445  36.227 165.623  38.291 175.397  44.012 183.301   44.37
 190.876  41.575 242.923  39.596
#Mann= 3 , 0 , 0
       0    .035       0       0    .035       0 242.923    .035       0
Bank Sta=0,242.923
XS Rating Curve= 0
Exp/Cntr=.3,.1

Type RM Length L Ch R = 1 ,772     ,59.055,59.055,59.055
XS GIS Cut Line= 2
      5314030.94     15922798.72      5313892.55     15923087.04
#Sta/Elev= 24
       0  54.173  30.574  53.054  43.714  43.159  49.928  42.812  55.515  39.134
  59.918  37.297  76.444  36.581  81.286  36.381  92.579  32.467 100.778  31.844
 113.668  31.627 123.176  30.994 136.713  31.552 147.523  30.833 154.006  31.962
 157.871  32.198 166.952  37.372 171.624  37.434 188.068  37.651 201.982  44.209
 212.966  44.459 257.375  44.475 285.197  52.831 320.597  53.648
#Mann= 3 , 0 , 0
       0    .035       0       0    .035       0 320.597    .035       0
Bank Sta=0,320.597
XS Rating Curve= 0
Exp/Cntr=.3,.1

Type RM Length L Ch R = 3 ,771.5   ,,,
BEGIN DESCRIPTION:
Bretellina
END DESCRIPTION:
Bridge Culvert--1,0,-1,-1, 0
Deck Dist Width WeirC Skew NumUp NumDn MinLoCord MaxHiCord MaxSubmerge Is_Ogee
1.64,55.774,2.61,0, 30, 30, , , .95, 0, 0,0,,
       0  30.545  43.701  43.701  49.869  55.479  59.744   78.74   78.74  81.168
  81.168  92.388 100.525 113.386   122.9  136.45 147.244 153.707 157.513 166.339
 166.339 168.963 168.963 187.533 201.411 212.336 256.693 256.693 284.416 319.783
  61.778  61.778  61.778  61.778  61.778  61.778  61.778  61.778  61.778  61.778
  61.778  61.778  61.778  61.778  61.778  61.778  61.778  61.778  61.778  61.778
  61.778  61.778  61.778  61.778  61.778  61.778  61.778  61.778  61.778  61.778
  54.167  53.051  43.143  50.131  50.131  50.131  50.131  50.131  36.319  36.352
  50.131  50.131  50.131  50.131  50.131  50.131  50.131  50.131  50.131  50.131
  37.467  37.402  50.131  50.131  50.131  50.131  49.869  44.488  50.131  50.131
       0  30.545  43.701  43.701  49.869  55.479  59.744   78.74   78.74  81.168
  81.168  92.388 100.525 113.386   122.9  136.45 147.244 153.707 157.513 166.339
 166.339 168.963 168.963 187.533 201.411 212.336 256.693 256.693 284.416 319.783
  61.778  61.778  61.778  61.778  61.778  61.778  61.778  61.778  61.778  61.778
  61.778  61.778  61.778  61.778  61.778  61.778  61.778  61.778  61.778  61.778
  61.778  61.778  61.778  61.778  61.778  61.778  61.778  61.778  61.778  61.778
  54.167  53.051  43.143  50.131  50.131  50.131  50.131  50.131  36.319  36.352
  50.131  50.131  50.131  50.131  50.131  50.131  50.131  50.131  50.131  50.131
  37.467  37.402  50.131  50.131  50.131  50.131  49.869  44.488  50.131  50.131
BR Coef=-1 , 0 , 0 ,1.25, 0 ,,,.8,-1,2,0,
WSPro=,,,, 1 ,,,, 0 ,,,, 0 ,,,,-1 ,-1 ,-1 , 0 , 0 , 0 , 0 , 0
BC Design=,, 0 ,, 0 ,,,,,,
BC HTab Sub Flow Pts= 40

Type RM Length L Ch R = 1 ,771.3   ,8.333,8.333,8.333
XS GIS Cut Line= 2
      5314030.94     15922798.72      5313892.55     15923087.04
#Sta/Elev= 24
       0  54.173  30.574  53.054  43.714  43.159  49.928  42.812  55.515  39.134
  59.918  37.297  76.444  36.581  81.286  36.381  92.579  32.467 100.778  31.844
 113.668  31.627 123.176  30.994 136.713  31.552 147.523  30.833 154.006  31.962
 157.871  32.198 166.952  37.372 171.624  37.434 188.068  37.651 201.982  44.209
 212.966  44.459 257.375  44.475 285.197  52.831 320.597  53.648
#Mann= 3 , 0 , 0
       0    .035       0       0    .035       0 320.597    .035       0
Bank Sta=0,320.597
XS Rating Curve= 0
Exp/Cntr=.3,.1

Type RM Length L Ch R = 1 ,771     ,76.936,76.936,76.936
XS GIS Cut Line= 2
       5313985.2     15922794.42       5313860.4      15923070.6
#Sta/Elev= 30
       0  55.148    8.77  54.738   10.81  51.722  12.493  51.355  15.925  53.891
  24.885  48.615  29.081  45.151  32.441  44.003    53.1  42.448  59.137  38.314
  72.694  38.363  75.814   37.27   82.31  36.742  90.259  36.476  100.84  34.882
   107.7  31.644 119.721  31.486 131.453  31.243 144.767  31.243 160.801   30.82
 174.131  30.075 180.889  30.249 187.359  30.459 196.726  37.192 211.083  37.372
 224.911  43.842 243.104  44.147 256.253  51.729 287.008   53.78 310.499  53.504
#Mann= 3 , 0 , 0
       0    .035       0       0    .035       0 310.499    .035       0
Bank Sta=0,310.499
XS Rating Curve= 0
Exp/Cntr=.3,.1

Type RM Length L Ch R = 1 ,770     ,168.898,168.898,168.898
XS GIS Cut Line= 2
      5313779.49     15922850.39      5313910.66     15923059.74
#Sta/Elev= 22
       0  41.516  28.143  41.985  37.497  46.122  57.536  46.739   82.94  36.581
  93.406  36.027 102.677  32.405 103.314  31.611 107.228   31.27 117.405  30.262
 127.674  31.211   137.9  30.912 148.789   31.43 153.832  31.519 160.965  36.663
 171.007   37.07 179.892  42.838 188.583  43.104  201.85  52.592 207.011  53.802
 230.538  53.671   247.5  53.041
#Mann= 3 , 0 , 0
       0    .035       0       0    .035       0   247.5    .035       0
Bank Sta=0,247.5
XS Rating Curve= 0
Exp/Cntr=.3,.1

Type RM Length L Ch R = 1 ,769     ,97.113,97.113,97.113
XS GIS Cut Line= 2
      5313634.38     15923005.38      5313851.97     15923174.77
#Sta/Elev= 27
       0  41.102   24.36   40.86  39.672  48.661  42.631  49.327  56.962   49.15
  61.001  48.205  82.182  37.428  98.196  35.689 102.421  32.907 102.818  31.995
 108.888  30.942 116.424  30.919 126.893  30.531 139.751  31.234 148.812  31.568
 153.743  31.594 158.783  31.814 167.313  35.735 181.939  37.372 192.106  42.759
  205.63  42.497 208.944  40.643 211.079  40.633 212.149  41.572 215.377  41.601
 235.692  53.675 276.345  53.363
#Mann= 3 , 0 , 0
       0    .035       0       0    .035       0 276.345    .035       0
Bank Sta=0,276.345
XS Rating Curve= 0
Exp/Cntr=.3,.1

Type RM Length L Ch R = 6 ,768.55  ,,,
Lateral Weir Pos= 0
Lateral Weir End=                ,                ,        ,c10
Lateral Weir Distance=3.281
Lateral Weir WD=9.843
Lateral Weir Coef=3.01
Lateral Weir Is Ogee= 0
Lateral Weir WSCriteria=-1
Lateral Weir SE= 6
       0   49.21    3.28   49.21    3.28   40.33    68.9   40.33    68.9   49.21
      72   49.21

Type RM Length L Ch R = 1 ,768     ,158.629,158.629,158.629
XS GIS Cut Line= 3
      5313589.63     15923090.91      5313809.45     15923261.98
      5313809.48     15923262.01
#Sta/Elev= 23
       0   40.61  23.314  40.466  41.417  40.253  74.472  40.535  76.089  34.564
   83.96  31.102  90.886  31.919  106.06  30.892 115.459  30.892 124.888  31.017
 131.775  31.916 140.676  31.965 149.098  35.653 162.835  36.995 174.833   42.51
 194.833  43.392 208.199  41.398 210.167  39.839 212.539  39.849 214.203  41.496
 217.795  41.847  238.31  54.078 280.052  53.865
#Mann= 3 , 0 , 0
       0    .035       0       0    .035       0 280.052    .035       0
Bank Sta=0,280.052
XS Rating Curve= 0
Exp/Cntr=.3,.1

Type RM Length L Ch R = 1 ,767     ,175.098,175.098,175.098
XS GIS Cut Line= 3
       5313489.6     15923215.12      5313683.17     15923375.98
      5313683.17     15923375.98
#Sta/Elev= 25
       0  41.411  20.797  42.293   28.94  48.825  40.663  48.698  64.413  36.627
  79.058   35.39  85.292  32.851  91.883  30.919 102.119  30.942 113.379   30.24
 123.602  30.282 132.103   30.42 136.106  31.952 141.391  32.228 148.301  35.896
 160.167  36.394  172.09   42.94 184.085  42.976 192.969  39.879 227.864  41.467
 240.922  41.017 243.173  39.383 244.967  39.429 246.568  41.066  252.47  41.594
#Mann= 3 , 0 , 0
       0    .035       0       0    .035       0  252.47    .035       0
Bank Sta=0,252.47
XS Rating Curve= 0
Exp/Cntr=.3,.1

Type RM Length L Ch R = 1 ,766     ,160.4,160.4,160.4
XS GIS Cut Line= 2
      5313369.62     15923340.94      5313558.23      15923499.7
#Sta/Elev= 21
       0  41.982  28.783  42.044  40.246  47.799  54.633  48.238  79.052  36.539
  90.804  36.017  99.974  32.913 100.994  31.962 106.913  30.305 116.204  30.279
 124.888  30.249 136.978  30.594 148.261  31.266 152.812  31.611 158.927  34.688
 173.757  36.119 187.011  43.163 199.255  43.169 205.636  40.417 226.608  40.246
 247.011  39.951
#Mann= 3 , 0 , 0
       0    .035       0       0    .035       0 247.011    .035       0
Bank Sta=0,247.011
XS Rating Curve= 0
Exp/Cntr=.3,.1

Type RM Length L Ch R = 1 ,765     ,276.214,276.214,276.214
XS GIS Cut Line= 2
      5313268.21     15923457.02       5313408.5     15923584.97
#Sta/Elev= 20
       0  41.237  13.107  41.345  25.741  47.559  40.062  47.559  65.561  36.552
  80.141  34.682  85.016  33.182  85.728   31.43  90.676  31.194 101.782  30.338
 112.969  30.069 119.232  29.915 128.228  30.755 135.643  31.611 139.534  31.217
 145.384  34.501 160.289  36.014 172.028  42.835 184.954  42.835 190.056  41.302
#Mann= 3 , 0 , 0
       0    .035       0       0    .035       0 190.056    .035       0
Bank Sta=0,190.056
XS Rating Curve= 0
Exp/Cntr=.3,.1

Type RM Length L Ch R = 6 ,764.55  ,,,
Lateral Weir Pos= 3
Lateral Weir End=                ,                ,        ,c09
Lateral Weir Distance=3.281
Lateral Weir WD=9.843
Lateral Weir Coef=3.01
Lateral Weir Is Ogee= 0
Lateral Weir WSCriteria=-1
Lateral Weir SE= 6
       0   49.21    3.28   49.21    3.28   41.97  167.25   41.97  167.25   49.21
   171.5   49.21

Type RM Length L Ch R = 1 ,764     ,65.354,65.354,65.354
XS GIS Cut Line= 3
      5313100.26     15923608.17      5313181.43     15923776.87
      5313201.48      15923818.5
#Sta/Elev= 24
       0  39.813  11.257  40.413  28.448  51.906  61.575  51.381  95.095  37.064
 106.447  36.089 117.989  32.484 118.757   31.07 123.291  31.243 134.259  30.571
 145.443  30.682 153.107  29.265 160.997  31.591 164.239  31.841 170.325  31.995
 185.896  32.562 194.291  32.694 194.537   42.31 204.738  42.323 205.348  33.346
 211.165  33.228 214.603  40.509 218.163  42.434 236.266  42.073
#Mann= 3 , 0 , 0
       0    .035       0       0    .035       0 236.266    .035       0
Bank Sta=0,236.266
XS Rating Curve= 0
Exp/Cntr=.3,.1

Type RM Length L Ch R = 1 ,763     ,185.728,185.728,185.728
XS GIS Cut Line= 2
      5313085.63     15923612.66      5313105.09     15923830.45
#Sta/Elev= 22
       0  39.347   9.055  39.623  27.123  51.463  60.653  52.129  93.474  37.041
 107.536  35.797 116.732  33.077 117.726  32.418 123.504  31.286 131.404  30.594
 140.276  30.262 147.139  29.281  152.07  30.331  163.52  31.847  182.74  32.215
 191.722  30.669 191.906    43.1 203.143  42.723 204.019  41.703 207.566  41.463
 207.999  32.592 221.214  32.644
#Mann= 3 , 0 , 0
       0    .035       0       0    .035       0 221.214    .035       0
Bank Sta=0,221.214
XS Rating Curve= 0
Exp/Cntr=.3,.1

Type RM Length L Ch R = 1 ,762     ,77.592,77.592,77.592
XS GIS Cut Line= 3
      5312924.41     15923661.98      5312907.61      15923866.5
      5312907.61      15923866.5
#Sta/Elev= 23
       0  33.868  17.461  33.845  18.278  39.928  20.689  40.118  21.237  43.035
  25.341  43.271  25.974  45.243  27.598  45.118  27.772  32.297  43.274  31.703
  51.033  31.001  55.689  31.247  66.427  31.257  79.373  30.413  89.508  29.921
 101.329  30.942 106.447  32.228 111.122  35.633 125.141  36.644 136.512  42.159
  151.02  42.585 156.598  41.329 206.572  39.596
#Mann= 3 , 0 , 0
       0    .035       0       0    .035       0 206.572    .035       0
Bank Sta=0,206.572
XS Rating Curve= 0
Exp/Cntr=.3,.1

Type RM Length L Ch R = 1 ,761     ,145.538,145.538,145.538
XS GIS Cut Line= 3
      5312836.88     15923674.93      5312860.73     15923898.46
      5312860.73     15923898.46
#Sta/Elev= 18
       0  37.546  12.638  36.998   28.94   35.81  36.588  33.071  37.503  32.339
  42.943  31.594  51.949  30.919  60.997  29.281  74.193  30.587  81.332   31.27
  86.414  31.972   94.59  36.188 107.011   36.89 119.236  42.559  141.46  42.034
 145.886  39.593 197.949  38.678  226.23  38.684
#Mann= 3 , 0 , 0
       0    .035       0       0    .035       0  226.23    .035       0
Bank Sta=0,226.23
XS Rating Curve= 0
Exp/Cntr=.3,.1

Type RM Length L Ch R = 1 ,760     ,152.034,152.034,152.034
XS GIS Cut Line= 3
      5312656.76     15923717.85      5312794.06     15923950.92
      5312794.06     15923950.92
#Sta/Elev= 22
       0  42.953   5.653  46.115  30.925  45.495  45.919  37.218  61.896  35.771
  65.709  33.468  66.765  32.162  72.746  30.965  80.495  29.639  88.573  29.964
  98.235  30.942 105.279  31.283 112.592  31.972 116.847  32.211 124.268  35.945
  137.69  36.588 151.969  43.481 168.202  43.973 177.008  41.142 208.514  40.095
 241.785  39.823 273.425  39.705
#Mann= 3 , 0 , 0
       0    .035       0       0    .035       0 273.425    .035       0
Bank Sta=0,273.425
XS Rating Curve= 0
Exp/Cntr=.3,.1

Type RM Length L Ch R = 1 ,693     ,43.504,43.504,43.504
XS GIS Cut Line= 2
      5312529.86     15923779.89      5312632.02     15923980.41
#Sta/Elev= 18
       0  42.815  39.108  46.457  49.081  44.324  61.319  38.156  77.362  36.483
  84.219  33.661  85.827  31.562  93.077  29.823 107.251  28.543 126.608   29.79
 135.007  31.693 136.155  33.957  138.78  35.433 152.625  36.483 166.503  43.307
 183.891   44.16 190.157  40.715 225.066  40.125
#Mann= 3 , 0 , 0
       0    .035       0       0    .035       0 225.066    .035       0
Bank Sta=0,225.066
XS Rating Curve= 0
Exp/Cntr=.3,.1

Type RM Length L Ch R = 1 ,692     ,38.287,38.287,38.287
XS GIS Cut Line= 2
      5312515.09      15923791.4       5312564.7      15924006.3
#Sta/Elev= 17
       0  43.635  35.072  45.407  50.919  39.042  66.207  36.778  73.425   33.76
  74.639  31.726  79.888   29.79 100.098  28.543 118.176  29.954 125.591  31.594
 127.231  33.104  130.61    35.4 145.112  36.581 159.449  43.701 178.904  43.241
 185.236  40.322 220.538  39.797
#Mann= 3 , 0 , 0
       0    .035       0       0    .035       0 220.538    .035       0
Bank Sta=0,220.538
XS Rating Curve= 0
Exp/Cntr=.3,.1

Type RM Length L Ch R = 1 ,691     ,85.269,85.269,85.269
XS GIS Cut Line= 2
      5312504.56     15923801.77      5312539.93     15924025.26
#Sta/Elev= 19
       0  43.602  32.808   45.44  47.178  39.436  63.944  37.303  73.163  33.136
  74.213  31.955  82.579  29.495  83.858   29.79  84.154  29.954 103.707  28.576
 120.636  30.052 121.916  29.724 127.953  31.988  132.48  35.696 145.801  36.614
 158.235  42.454  182.48  43.209 186.909  41.175  226.28  41.043
#Mann= 3 , 0 , 0
       0    .035       0       0    .035       0  226.28    .035       0
Bank Sta=0,226.28
XS Rating Curve= 0
Exp/Cntr=.3,.1

Type RM Length L Ch R = 1 ,690     ,70.112,70.112,70.112
XS GIS Cut Line= 2
      5312467.91     15923741.27      5312380.77     15923968.21
#Sta/Elev= 18
       0  39.797  46.654  43.471  53.707  45.801  67.224  45.768  83.661  38.812
  94.291  37.959 102.034  35.958 102.854  31.529  109.35  29.462 129.593   28.74
 158.694  28.839 166.404  31.398 167.552  32.579 172.014  34.318 184.088  41.634
 204.888  41.306 208.694  39.797 243.077  39.239
#Mann= 3 , 0 , 0
       0    .035       0       0    .035       0 243.077    .035       0
Bank Sta=0,243.077
XS Rating Curve= 0
Exp/Cntr=.3,.1

Type RM Length L Ch R = 1 ,689     ,96.785,96.785,96.785
XS GIS Cut Line= 2
      5312412.89     15923730.09      5312300.98     15923940.55
#Sta/Elev= 21
       0  39.895   38.55  41.535  45.669   45.21  55.807  45.276   69.98   38.32
  90.322  35.991  91.043  33.694  92.749  33.596  94.259   31.43 101.181  29.626
 119.357  28.871 135.761  28.871 143.832  29.593 148.589  32.087 151.804  34.285
 161.089  39.731 167.323  40.748  178.15  41.896 190.682  42.028 195.702  40.551
 238.353  39.534
#Mann= 3 , 0 , 0
       0    .035       0       0    .035       0 238.353    .035       0
Bank Sta=0,238.353
XS Rating Curve= 0
Exp/Cntr=.3,.1

Type RM Length L Ch R = 1 ,688     ,87.205,87.205,87.205
XS GIS Cut Line= 2
      5312309.84     15923682.38      5312228.44     15923906.04
#Sta/Elev= 19
       0  41.765  48.819  43.045  50.951  44.554  57.907  43.996  71.522  37.959
  85.269  36.253   92.06  33.399  93.077  31.135  104.56  29.856 124.114  29.035
 138.747  28.937 146.555   31.43 147.539  33.268 163.156  40.157  178.51  41.043
 183.497   42.52 196.391  41.371 203.018  38.878 237.992  39.469
#Mann= 3 , 0 , 0
       0    .035       0       0    .035       0 237.992    .035       0
Bank Sta=0,237.992
XS Rating Curve= 0
Exp/Cntr=.3,.1

Type RM Length L Ch R = 1 ,687     ,83.235,83.235,83.235
XS GIS Cut Line= 2
      5312221.33     15923638.68      5312161.09     15923863.42
#Sta/Elev= 19
       0  40.814  51.345  42.552  56.266  44.915  65.223  43.734  76.772  37.566
  89.009  36.844  97.507  33.596  99.114  31.791 110.138  30.085 131.168  29.199
 144.193  29.035   152.1  31.529 156.299  34.088  164.14  38.123 184.678  40.617
 187.139  41.535 198.589  41.765 201.608   40.65 232.677  39.469
#Mann= 3 , 0 , 0
       0    .035       0       0    .035       0 232.677    .035       0
Bank Sta=0,232.677
XS Rating Curve= 0
Exp/Cntr=.3,.1

Type RM Length L Ch R = 1 ,686     ,72.113,72.113,72.113
XS GIS Cut Line= 2
      5312142.72     15923621.26      5312080.22     15923839.17
#Sta/Elev= 20
       0  41.142  33.235   42.06  40.715  45.243  48.097  44.587  59.843  38.091
  74.475  37.402  81.266  34.449  83.563  31.594  94.291  30.282 116.667  29.364
 128.215  29.101 137.959   31.89  139.14  33.169 152.789  38.812 166.601  39.993
 173.556  42.126 182.021  41.962 187.434  41.076 191.634  39.469 226.706  39.633
#Mann= 3 , 0 , 0
       0    .035       0       0    .035       0 226.706    .035       0
Bank Sta=0,226.706
XS Rating Curve= 0
Exp/Cntr=.3,.1

Type RM Length L Ch R = 1 ,685     ,65.026,65.026,65.026
XS GIS Cut Line= 2
      5312081.43     15923595.73      5312011.88      15923797.7
#Sta/Elev= 24
       0  40.879  30.741  41.404   34.81  44.324  44.455  44.324  53.117  38.615
  71.916  37.894  79.528  34.678  82.152  31.824  92.881  30.052  104.79  29.659
  110.86  30.446 116.273  29.495 131.365  29.167 135.663  29.626 139.206  31.496
 139.633  32.874 141.404  33.465 150.558    39.6  158.76  39.304 165.846  40.354
  169.98  41.601 184.088  41.175 191.699  39.337 213.615  38.615
#Mann= 3 , 0 , 0
       0    .035       0       0    .035       0 213.615    .035       0
Bank Sta=0,213.615
XS Rating Curve= 0
Exp/Cntr=.3,.1

Type RM Length L Ch R = 1 ,684     ,11.22,11.22,11.22
XS GIS Cut Line= 2
      5312036.09     15923577.66      5311938.88     15923768.44
#Sta/Elev= 15
       0  40.912      25  41.798  29.429  43.176  53.412  41.568  69.455  38.583
  80.217  33.858  82.021  31.857 110.433  28.937 116.142  29.593 133.399  29.199
 139.961  32.087 149.049  38.189 160.072  39.829 170.013  42.028 214.108  40.715
#Mann= 3 , 0 , 0
       0    .035       0       0    .035       0 214.108    .035       0
Bank Sta=0,214.108
XS Rating Curve= 0
Exp/Cntr=.3,.1

Type RM Length L Ch R = 1 ,683.2   ,22.966,22.966,22.966
XS GIS Cut Line= 2
      5312024.11     15923550.85      5311964.63     15923698.06
#Sta/Elev= 15
       0  41.207  24.573  41.142  29.003   42.52  53.412  41.568  69.455  38.583
  80.315  33.333 110.433  33.333  113.32  33.333  121.85  28.084 133.005  28.543
 139.961  32.119 149.049  38.189 160.072  39.895 170.013  42.028 214.108  40.748
#Mann= 3 , 0 , 0
       0    .035       0       0    .035       0 214.108    .035       0
Bank Sta=0,214.108
XS Rating Curve= 0
Exp/Cntr=.3,.1

Type RM Length L Ch R = 3 ,683.1   ,,,
BEGIN DESCRIPTION:
Cateratte
END DESCRIPTION:
Bridge Culvert--1,0,-1,-1, 0
Deck Dist Width WeirC Skew NumUp NumDn MinLoCord MaxHiCord MaxSubmerge Is_Ogee
1.64,19.685,2.61,0, 27, 27, , , .95, 0, 0,0,,
  29.003  53.412  80.315  80.315   88.78   88.78  91.142  91.142  99.475  99.475
 101.772 101.772 110.433 110.433  113.32  113.32  121.85  121.85 124.967 124.967
 133.005 133.005 139.961 149.049 160.072 170.013 173.885
   42.52   42.52  43.176  43.176  43.176  43.176  43.176  43.176  43.176  43.176
  43.176  43.176  43.176  43.176  43.176  43.176  43.176  43.176  43.176  43.176
  43.176  43.176  43.176  43.176  43.176  43.176  41.896
   42.52  41.568  33.333  42.126  42.126  33.333  33.333  42.126  42.126  33.333
  33.333  42.126  42.126  33.333  33.333  42.126  42.126  28.084  28.281  42.126
  42.126  28.543  32.119  38.189  39.895  42.028  41.896
  29.003  53.412  80.315  80.315   88.78   88.78  91.142  91.142  99.475  99.475
 101.772 101.772 110.433 110.433  113.32  113.32  121.85  121.85 124.967 124.967
 133.005 133.005 139.961 149.049 160.072 170.013 173.885
   42.52   42.52  43.176  43.176  43.176  43.176  43.176  43.176  43.176  43.176
  43.176  43.176  43.176  43.176  43.176  43.176  43.176  43.176  43.176  43.176
  43.176  43.176  43.176  43.176  43.176  43.176  41.896
   42.52  41.568  33.333  42.126  42.126  33.333  33.333  42.126  42.126  33.333
  33.333  42.126  42.126  33.333  33.333  42.126  42.126  28.084  28.281  42.126
  42.126  28.543  32.119  38.189  39.895  42.028  41.896
BR Coef=-1 , 0 , 0 ,1.25, 0 ,,,.8,-1,2,0,
WSPro=,,,, 1 ,,,, 0 ,,,, 0 ,,,,-1 ,-1 ,-1 , 0 , 0 , 0 , 0 , 0
BC Design=,, 0 ,, 0 ,,,,,,
BC HTab Sub Flow Pts= 40

Type RM Length L Ch R = 1 ,683     ,6.234,6.234,6.234
XS GIS Cut Line= 2
      5312024.11     15923550.85      5311964.63     15923698.06
#Sta/Elev= 15
       0  41.207  24.573  41.142  29.003   42.52  53.412  41.568  69.455  38.583
  80.315  33.333 110.433  33.333  113.32  33.333  121.85  28.084 133.005  28.543
 139.961  32.119 149.049  38.189 160.072  39.895 170.013  42.028 214.108  40.748
#Mann= 3 , 0 , 0
       0    .035       0       0    .035       0 214.108    .035       0
Bank Sta=0,214.108
XS Rating Curve= 0
Exp/Cntr=.3,.1

Type RM Length L Ch R = 1 ,682     ,128.576,128.576,128.576
XS GIS Cut Line= 2
      5311900.46     15923561.29      5311951.35     15923781.66
#Sta/Elev= 15
       0  40.814   25.82  42.323  39.961  41.568  55.774  35.007  57.021  34.154
  66.864   31.66 102.428  30.741 112.008  28.839 129.068  28.346 139.075  31.726
 141.699  33.694 154.954  41.765 182.283  42.388 183.465  41.798 226.181  40.715
#Mann= 3 , 0 , 0
       0    .035       0       0    .035       0 226.181    .035       0
Bank Sta=0,226.181
XS Rating Curve= 0
Exp/Cntr=.3,.1

Type RM Length L Ch R = 1 ,681     ,82.448,82.448,82.448
XS GIS Cut Line= 2
      5311758.76     15923613.45       5311904.3     15923786.88
#Sta/Elev= 18
       0  40.617   34.35  41.306  42.618  41.962  46.916  40.289  50.591   37.27
  60.072  36.713  65.125  31.791  72.014  28.839  92.585  29.626   110.4  28.445
 119.324  31.791 121.129  34.843 128.543  37.762 146.883  39.239 153.478  41.864
 171.063  42.224 180.151  42.454 226.411   40.65
#Mann= 3 , 0 , 0
       0    .035       0       0    .035       0 226.411    .035       0
Bank Sta=0,226.411
XS Rating Curve= 0
Exp/Cntr=.3,.1

Type RM Length L Ch R = 1 ,680     ,94.455,94.455,94.455
XS GIS Cut Line= 2
      5311697.24     15923675.39      5311843.34     15923832.09
#Sta/Elev= 21
       0  40.223  30.249  40.879  34.744  42.323   40.19  42.323  46.719  39.698
  49.016  35.531  63.845   34.81  66.601  31.004  73.163  28.904  90.748  29.232
 104.724  28.609  109.58  31.955 110.794  33.333 116.962  36.713 130.315   37.73
 149.573  40.518 152.789  38.747  161.45  39.567 166.109  41.831 176.444  41.995
 214.239  41.273
#Mann= 3 , 0 , 0
       0    .035       0       0    .035       0 214.239    .035       0
Bank Sta=0,214.239
XS Rating Curve= 0
Exp/Cntr=.3,.1

Type RM Length L Ch R = 1 ,679     ,74.213,74.213,74.213
XS GIS Cut Line= 2
      5311630.41     15923734.88      5311770.18     15923901.41
#Sta/Elev= 20
       0  40.026  35.302  40.781  39.534  42.585  49.344  42.421   54.79  39.993
  57.251  36.417  69.324  35.203  72.047  31.529  81.102   28.97  95.702  28.773
 106.955  28.806 118.209  31.857 122.933  35.892 140.092  38.615 152.592  39.534
 157.612  38.747 166.995  39.403  173.95  41.601 184.383  42.028 217.421  41.765
#Mann= 3 , 0 , 0
       0    .035       0       0    .035       0 217.421    .035       0
Bank Sta=0,217.421
XS Rating Curve= 0
Exp/Cntr=.3,.1

Type RM Length L Ch R = 1 ,678     ,73.983,73.983,73.983
XS GIS Cut Line= 2
      5311582.91      15923776.9      5311695.41      15923943.7
#Sta/Elev= 21
       0  40.256  30.676  40.978  35.663  42.618  43.799  42.224  43.963  42.192
  54.659  37.434  71.621  35.761  77.854  31.529  88.517  29.035 101.017  28.412
 110.236  28.937 124.278  31.988 125.295  33.071 130.348  36.286 141.601  37.598
 146.227  39.173 160.794  41.896 162.467  41.076 166.732   40.65 170.571  41.864
 201.181  41.864
#Mann= 3 , 0 , 0
       0    .035       0       0    .035       0 201.181    .035       0
Bank Sta=0,201.181
XS Rating Curve= 0
Exp/Cntr=.3,.1

Type RM Length L Ch R = 1 ,677     ,88.747,88.747,88.747
XS GIS Cut Line= 2
      5311513.98     15923810.43      5311629.86     15923975.95
#Sta/Elev= 18
       0  39.961  37.008  41.076  40.223  42.684  49.213  42.881  55.479  39.567
  66.929  37.402  78.806  37.664  87.402  35.072  91.995  31.955  96.457  29.068
 116.273  28.117 128.215  27.854 140.322  32.054 142.913  34.711 145.866   35.63
  175.82  37.303 190.912  41.535 202.067  41.864
#Mann= 3 , 0 , 0
       0    .035       0       0    .035       0 202.067    .035       0
Bank Sta=0,202.067
XS Rating Curve= 0
Exp/Cntr=.3,.1

Type RM Length L Ch R = 1 ,676     ,78.871,78.871,78.871
XS GIS Cut Line= 2
       5311441.6     15923850.79      5311573.36     15924061.61
#Sta/Elev= 17
       0  39.829  39.009  40.814  41.535  42.192  54.724   42.06  60.958  38.845
  86.811  37.697  92.356  36.089  98.917  31.791 102.362  29.724 120.702  28.609
 135.007  27.723  147.08  31.791 151.509  36.188 178.576  35.827 195.308  41.535
 208.891  41.634 248.622  41.273
#Mann= 3 , 0 , 0
       0    .035       0       0    .035       0 248.622    .035       0
Bank Sta=0,248.622
XS Rating Curve= 0
Exp/Cntr=.3,.1

Type RM Length L Ch R = 1 ,675     ,91.404,91.404,91.404
XS GIS Cut Line= 2
      5311376.54     15923891.57      5311513.06     15924118.77
#Sta/Elev= 19
       0    39.6   37.27  40.289  40.748   42.06  49.213   42.06  55.249  39.829
  84.121  36.516  87.631  35.302   93.57  31.726  100.82  30.348 101.608  30.381
 119.685  29.134 135.171  27.592 142.585  31.332 150.459  35.958 183.301  37.073
 192.224  41.864 205.938  41.929 208.465  39.961 265.059  41.634
#Mann= 3 , 0 , 0
       0    .035       0       0    .035       0 265.059    .035       0
Bank Sta=0,265.059
XS Rating Curve= 0
Exp/Cntr=.3,.1

Type RM Length L Ch R = 1 ,674     ,93.602,93.602,93.602
XS GIS Cut Line= 2
       5311306.5     15923941.04      5311423.13     15924160.43
#Sta/Elev= 18
       0  39.436  29.528  39.797  34.383  42.651  44.029  41.995  51.444  39.173
  71.686  36.417  76.444  33.465  79.593  31.529  87.238  29.823 105.873  29.003
 123.589  28.445 135.564  32.021 139.206  34.875 174.541  37.992 181.726  41.175
 196.752   41.24 199.541  39.469 248.458  40.486
#Mann= 3 , 0 , 0
       0    .035       0       0    .035       0 248.458    .035       0
Bank Sta=0,248.458
XS Rating Curve= 0
Exp/Cntr=.3,.1

Type RM Length L Ch R = 1 ,673     ,93.307,93.307,93.307
XS GIS Cut Line= 2
      5311236.52     15923972.18      5311317.06      15924206.1
#Sta/Elev= 20
       0   40.19  37.533  40.912  41.437  42.585  53.576  42.126   58.76  38.419
  69.357  37.664  79.659  31.332  89.797  29.298 109.383  28.839 129.757  29.331
 139.042  31.562 142.224  33.136 144.915  35.925 162.697  35.958 167.946  37.369
 178.182  38.123 183.301  41.634 195.965  41.995     200  38.845 247.408  39.337
#Mann= 3 , 0 , 0
       0    .035       0       0    .035       0 247.408    .035       0
Bank Sta=0,247.408
XS Rating Curve= 0
Exp/Cntr=.3,.1

Type RM Length L Ch R = 1 ,672     ,49.803,49.803,49.803
XS GIS Cut Line= 2
      5311139.93     15923983.89      5311214.11      15924187.7
#Sta/Elev= 16
       0  40.092  32.513  40.682  47.572  42.815  75.984  41.896  76.017  41.864
   90.19  33.136  95.079   31.89 103.412  29.298 120.866  28.839 142.717  29.331
 150.755  32.251 153.543  33.497 155.577  35.433 170.177  41.896 203.248  41.568
 216.896  38.583
#Mann= 3 , 0 , 0
       0    .035       0       0    .035       0 216.896    .035       0
Bank Sta=0,216.896
XS Rating Curve= 0
Exp/Cntr=.3,.1

Type RM Length L Ch R = 1 ,671.5   ,32.808,32.808,32.808
#Sta/Elev= 16
       0  45.112  63.911  43.077  80.217  44.029  92.585  41.371  99.311  31.824
 110.499  29.396 111.844  29.396 113.353  29.364 127.198  29.298 141.273  29.528
 142.782   29.56 148.786  29.659 158.136  32.087 161.417  34.186 177.165  43.701
 201.444  43.471
#Mann= 3 , 0 , 0
       0    .035       0       0    .035       0 201.444    .035       0
Bank Sta=0,201.444
XS Rating Curve= 0
Exp/Cntr=.3,.1

Type RM Length L Ch R = 3 ,671.3   ,,,
BEGIN DESCRIPTION:
Ponte di ferro
END DESCRIPTION:
Bridge Culvert--1,0,-1,-1, 0
Deck Dist Width WeirC Skew NumUp NumDn MinLoCord MaxHiCord MaxSubmerge Is_Ogee
1.64,29.528,2.61,0, 14, 14, , , .95, 0, 0,0,,
  80.217  92.585  92.585 111.844 111.844 113.353 113.353 141.273 141.273 142.782
 142.782 161.417 161.417 177.165
  44.029  44.029  44.029  44.029  44.029  44.029  44.029  44.029  44.029  44.029
  44.029  44.029  44.029  43.701
  44.029  34.908  42.126  42.126  29.396  29.364  42.126  42.126  29.528   29.56
  42.126  42.126  34.186  43.701
  80.217  92.585  92.585 111.844 111.844 113.353 113.353 141.273 141.273 142.782
 142.782 161.417 161.417 177.165
  44.029  44.029  44.029  44.029  44.029  44.029  44.029  44.029  44.029  44.029
  44.029  44.029  44.029  43.701
  44.029  34.908  42.126  42.126  29.396  29.364  42.126  42.126  29.528   29.56
  42.126  42.126  34.186  43.701
BR Coef=-1 , 0 , 0 ,1.25, 0 ,,,.8,-1,2,0,
WSPro=,,,, 1 ,,,, 0 ,,,, 0 ,,,,-1 ,-1 ,-1 , 0 , 0 , 0 , 0 , 0
BC Design=,, 0 ,, 0 ,,,,,,
BC HTab Sub Flow Pts= 40

Type RM Length L Ch R = 1 ,671.2   ,13.451,13.451,13.451
#Sta/Elev= 16
       0  45.112  63.911  43.077  80.217  44.029  92.585  41.371  99.311  31.824
 110.499  29.396 111.844  29.396 113.353  29.364 127.198  29.298 141.273  29.528
 142.782   29.56 148.786  29.659 158.136  32.087 161.417  34.186 177.165  43.701
 201.444  43.471
#Mann= 3 , 0 , 0
       0    .035       0       0    .035       0 201.444    .035       0
Bank Sta=0,201.444
XS Rating Curve= 0
Exp/Cntr=.3,.1

Type RM Length L Ch R = 1 ,671     ,90.551,90.551,90.551
XS GIS Cut Line= 2
      5311124.67     15923996.92      5311190.26     15924187.37
#Sta/Elev= 12
       0   44.16  63.944  42.126  75.295  36.286  80.741  32.054   94.16   29.79
 110.072  30.118  131.43  30.348 142.192  32.251 146.161  35.203 157.415  39.567
 162.106  42.979 201.444   42.52
#Mann= 3 , 0 , 0
       0    .035       0       0    .035       0 201.444    .035       0
Bank Sta=0,201.444
XS Rating Curve= 0
Exp/Cntr=.3,.1

Type RM Length L Ch R = 1 ,670     ,85.007,85.007,85.007
XS GIS Cut Line= 2
      5311049.67     15924014.11      5311094.98      15924227.2
#Sta/Elev= 20
       0  40.551  32.907   40.42  37.402   43.34  48.917  43.176  57.546   37.73
  83.661  36.122  85.761  34.875  87.828  31.562  89.862  29.495 104.659   29.79
 123.753   30.02 135.827   31.43 137.073  33.038  144.16  33.235 146.293    35.4
 154.265  36.155 161.877  42.717 177.034  42.913 181.168  40.945 217.848  39.961
#Mann= 3 , 0 , 0
       0    .035       0       0    .035       0 217.848    .035       0
Bank Sta=0,217.848
XS Rating Curve= 0
Exp/Cntr=.3,.1

Type RM Length L Ch R = 1 ,669     ,83.038,83.038,83.038
XS GIS Cut Line= 2
      5310964.99     15924013.85      5311009.42     15924242.32
#Sta/Elev= 20
       0  40.617  33.661  41.503  37.205  43.602  47.211  44.094  57.907  37.959
  90.978  37.106  99.049  33.629 100.886  31.463 103.707  29.134 119.029  28.806
 136.319  28.904 150.295  30.971 151.739  34.252 163.222  37.533 173.163   42.29
 185.105  43.045 191.076  37.303  193.11  37.369 195.965  38.911 232.743  39.469
#Mann= 3 , 0 , 0
       0    .035       0       0    .035       0 232.743    .035       0
Bank Sta=0,232.743
XS Rating Curve= 0
Exp/Cntr=.3,.1

Type RM Length L Ch R = 1 ,668     ,74.278,74.278,74.278
XS GIS Cut Line= 2
      5310886.48     15924021.78      5310923.95     15924258.17
#Sta/Elev= 21
       0  40.157  35.367  41.601  38.714  43.438  47.999  43.799  57.612  37.861
  86.713  37.336  101.05  34.514 102.822  31.726 108.825  28.904 124.738  28.314
  140.42  28.314 147.736  30.807 153.346  34.154 156.726  36.286 165.978  37.303
 175.295  42.717 189.436  42.454 196.982  37.959 199.213  37.959 200.689  39.272
 239.337  39.501
#Mann= 3 , 0 , 0
       0    .035       0       0    .035       0 239.337    .035       0
Bank Sta=0,239.337
XS Rating Curve= 0
Exp/Cntr=.3,.1

Type RM Length L Ch R = 1 ,667     ,86.024,86.024,86.024
XS GIS Cut Line= 2
       5310799.8     15924034.51      5310865.12     15924278.22
#Sta/Elev= 22
       0  40.092  44.915  41.306  49.541  43.077  53.314  43.373  57.382  43.012
  66.043  37.697 100.656  35.564 103.609  31.594 111.516   28.74  128.15  27.953
 143.373  27.887 150.787  31.791 152.526  33.727 159.613  37.041 174.803  38.451
 184.875  42.782 201.444  42.749 208.005  40.518 210.696  37.992 212.959  38.353
 214.797  39.567 252.297  39.633
#Mann= 3 , 0 , 0
       0    .035       0       0    .035       0 252.297    .035       0
Bank Sta=0,252.297
XS Rating Curve= 0
Exp/Cntr=.3,.1

Type RM Length L Ch R = 1 ,666     ,76.181,76.181,76.181
XS GIS Cut Line= 2
      5310701.21      15924104.1      5310823.72     15924308.01
#Sta/Elev= 20
       0   41.01  45.308   42.29  56.398  41.798  64.206   38.55   70.21  36.942
  77.264  31.102   82.94   28.51 102.526   28.74 120.669  28.609 126.837  31.562
 129.659  34.088 135.138  37.533 170.341  37.697 182.415  42.946 196.194   42.29
 200.558  40.617  203.15  37.927 204.692  37.927 206.463  38.714 237.861  39.928
#Mann= 3 , 0 , 0
       0    .035       0       0    .035       0 237.861    .035       0
Bank Sta=0,237.861
XS Rating Curve= 0
Exp/Cntr=.3,.1

Type RM Length L Ch R = 1 ,665     ,90.322,90.322,90.322
XS GIS Cut Line= 2
      5310634.48     15924146.92       5310750.2      15924325.1
#Sta/Elev= 16
       0  40.978  41.371  42.815    52.1  42.356  64.042  36.024  68.471  31.332
  79.495  28.773  92.651  28.576 111.581  28.543 116.798  31.955 120.997  36.745
 151.115  38.222 152.822  36.975 165.584  37.303 176.148  41.995 187.926  42.717
 212.467  43.668
#Mann= 3 , 0 , 0
       0    .035       0       0    .035       0 212.467    .035       0
Bank Sta=0,212.467
XS Rating Curve= 0
Exp/Cntr=.3,.1

Type RM Length L Ch R = 1 ,664     ,85.794,85.794,85.794
XS GIS Cut Line= 2
      5310557.45     15924205.64      5310692.26     15924384.55
#Sta/Elev= 15
       0  40.584  42.028  41.962  46.227  42.618  53.281   42.06  68.701  34.219
  70.571  31.398   81.07  29.035  97.146  28.412 106.463  28.478 117.749  31.562
 123.983  36.253 148.622  38.911 167.126  37.073 178.806  40.978 224.016  41.109
#Mann= 3 , 0 , 0
       0    .035       0       0    .035       0 224.016    .035       0
Bank Sta=0,224.016
XS Rating Curve= 0
Exp/Cntr=.3,.1

Type RM Length L Ch R = 1 ,663     ,82.48,82.48,82.48
XS GIS Cut Line= 2
      5310493.24     15924265.42      5310621.03     15924428.97
#Sta/Elev= 14
       0  40.814  39.993  42.454  44.652   42.29  58.891  35.564  62.073  31.463
   74.18  29.298  92.979  28.248 106.529  28.412 115.453  31.529 123.753  36.745
 162.598  37.434 172.605  41.109 178.806  41.634 207.546  40.617
#Mann= 3 , 0 , 0
       0    .035       0       0    .035       0 207.546    .035       0
Bank Sta=0,207.546
XS Rating Curve= 0
Exp/Cntr=.3,.1

Type RM Length L Ch R = 1 ,662     ,80.643,80.643,80.643
XS GIS Cut Line= 2
      5310422.15     15924311.12      5310566.04     15924488.81
#Sta/Elev= 15
       0  40.879  51.837  41.175  60.794  36.778  75.591  34.514  77.198  30.774
  82.218   29.56 103.839  28.084 121.686  28.346 126.706  31.332 133.301  36.024
 169.554  37.795 177.559  41.043 186.122  41.535 193.471  40.387 228.642  40.453
#Mann= 3 , 0 , 0
       0    .035       0       0    .035       0 228.642    .035       0
Bank Sta=0,228.642
XS Rating Curve= 0
Exp/Cntr=.3,.1

Type RM Length L Ch R = 1 ,661     ,87.5,87.5,87.5
XS GIS Cut Line= 2
      5310355.02     15924355.81      5310499.34     15924534.02
#Sta/Elev= 16
       0  40.486  59.285  41.404  72.014  37.631  88.583  35.105  92.913  31.037
  97.146  29.495  118.34  28.084 136.385  28.314 141.273  31.365 143.668  34.285
 151.312  36.778 179.757   39.14 184.547  40.846 198.163  41.306  207.48  40.092
 229.331  39.993
#Mann= 3 , 0 , 0
       0    .035       0       0    .035       0 229.331    .035       0
Bank Sta=0,229.331
XS Rating Curve= 0
Exp/Cntr=.3,.1

Type RM Length L Ch R = 1 ,660     ,81.529,81.529,81.529
XS GIS Cut Line= 2
      5310293.57     15924424.57      5310448.98     15924603.38
#Sta/Elev= 19
       0  40.157  46.325  41.437  55.479  41.109  61.581  38.681  74.278  37.795
  81.726  33.629  83.629  31.824  90.715  29.429 111.549  28.084  128.97  28.314
 132.612  31.857 138.451  36.024 147.572  37.369 159.744  36.713 170.702  37.106
 182.185  40.584 192.126  41.043 196.391  39.403 236.909    39.6
#Mann= 3 , 0 , 0
       0    .035       0       0    .035       0 236.909    .035       0
Bank Sta=0,236.909
XS Rating Curve= 0
Exp/Cntr=.3,.1

Type RM Length L Ch R = 1 ,659     ,85.531,85.531,85.531
XS GIS Cut Line= 2
      5310247.28     15924500.07      5310397.47     15924661.15
#Sta/Elev= 19
       0  39.928  29.987  40.551   42.06  41.142  46.227  39.173  50.787  38.189
  57.808  34.449  60.203  31.693  68.898  29.396  89.501  28.051 106.398  28.281
  110.86  31.857 113.878  34.186 124.114  36.319  148.72  36.188 159.514  36.286
 171.621  40.715 179.921  41.339 184.908  39.108 220.243  39.272
#Mann= 3 , 0 , 0
       0    .035       0       0    .035       0 220.243    .035       0
Bank Sta=0,220.243
XS Rating Curve= 0
Exp/Cntr=.3,.1

Type RM Length L Ch R = 1 ,658     ,93.668,93.668,93.668
XS GIS Cut Line= 2
      5310192.49     15924547.57      5310323.06     15924734.06
#Sta/Elev= 18
       0  39.403  34.121  41.142  47.671  40.879  55.709  36.811  64.042  35.203
  65.879  33.235  67.192  33.104  68.209  30.873  73.392  29.331  94.259  28.051
 111.056  28.248  121.26  31.562 124.508  34.383 131.791  36.286 151.476  36.417
 171.522  37.369 178.445  40.617 227.657  40.814
#Mann= 3 , 0 , 0
       0    .035       0       0    .035       0 227.657    .035       0
Bank Sta=0,227.657
XS Rating Curve= 0
Exp/Cntr=.3,.1

Type RM Length L Ch R = 1 ,657     ,80.184,80.184,80.184
XS GIS Cut Line= 2
      5310111.45     15924600.07      5310246.62     15924779.46
#Sta/Elev= 17
       0  39.862  33.891  40.453  47.474  41.175  56.529  37.106  74.114  36.188
  84.285  34.482  86.975  31.398  93.176  29.265 111.549  28.051 128.117  28.215
 136.352  30.906 138.255  33.924 148.327   36.22 162.074   37.27 171.522  41.568
 187.533  41.896 224.606  41.437
#Mann= 3 , 0 , 0
       0    .035       0       0    .035       0 224.606    .035       0
Bank Sta=0,224.606
XS Rating Curve= 0
Exp/Cntr=.3,.1

Type RM Length L Ch R = 1 ,656     ,116.404,116.404,116.404
XS GIS Cut Line= 2
      5310055.45     15924618.64      5310152.36     15924817.36
#Sta/Elev= 20
       0  39.928  39.764  40.486  40.715  41.273  53.773  40.879  60.466  37.434
  83.924  36.385  99.245  35.531 102.822  34.318 105.315   31.89 111.417  29.068
 122.638  28.117 138.386  28.182 151.837  31.234 155.151  35.236 168.668   36.68
 169.094  38.714 175.558  41.437 181.102  41.831 187.073  41.503 221.096  40.617
#Mann= 3 , 0 , 0
       0    .035       0       0    .035       0 221.096    .035       0
Bank Sta=0,221.096
XS Rating Curve= 0
Exp/Cntr=.3,.1

Type RM Length L Ch R = 1 ,655     ,87.762,87.762,87.762
XS GIS Cut Line= 2
      5309935.37     15924686.06      5310072.24     15924874.44
#Sta/Elev= 19
       0  39.501  38.287   40.19  41.076  41.175  52.034   41.01  56.693  38.451
  76.181  36.713  88.123  35.302  91.503  33.858  93.209  31.594 102.887   28.74
 124.049  28.084 138.976   28.15 148.031  31.529 153.215  35.892 164.272  36.647
 172.835  41.864 183.301  41.371 187.926  39.895 232.874  38.845
#Mann= 3 , 0 , 0
       0    .035       0       0    .035       0 232.874    .035       0
Bank Sta=0,232.874
XS Rating Curve= 0
Exp/Cntr=.3,.1

Type RM Length L Ch R = 1 ,654     ,116.667,116.667,116.667
XS GIS Cut Line= 2
       5309858.3     15924756.86       5310035.4     15924933.96
#Sta/Elev= 19
       0  39.337  40.026  41.535  51.115  41.306  60.499  36.516   78.74  35.335
  82.218  32.907  83.005  31.266  88.681  28.478 104.101   28.15 118.143  28.117
 129.921  31.529 131.594  33.005 135.007  35.007 164.337   36.45 173.852  41.732
 179.659  42.585 188.648   42.06 196.358  39.534 250.459  38.976
#Mann= 3 , 0 , 0
       0    .035       0       0    .035       0 250.459    .035       0
Bank Sta=0,250.459
XS Rating Curve= 0
Exp/Cntr=.3,.1
