HEC-RAS study ozz_def.prj: ozzeri

--- ozz_def.g04 (geometry) --- (continued)

Type RM Length L Ch R = 1 ,653     ,89.829,89.829,89.829
XS GIS Cut Line= 2
      5309780.31     15924886.55      5309997.24      15924987.7
#Sta/Elev= 17
       0   39.14  36.122  39.436  40.879  41.568  52.297  41.109  64.009    35.4
  68.241  31.791  78.675  29.593  95.177  27.428 108.858  26.706 113.091   31.43
  117.29  34.449 141.142  36.385 164.633  36.942 174.278  41.634 185.761   42.06
 195.079  39.633 239.337  38.878
#Mann= 3 , 0 , 0
       0    .035       0       0    .035       0 239.337    .035       0
Bank Sta=0,239.337
XS Rating Curve= 0
Exp/Cntr=.3,.1

Type RM Length L Ch R = 1 ,652     ,71.063,71.063,71.063
XS GIS Cut Line= 2
      5309744.32     15924972.38      5309946.92     15925058.37
#Sta/Elev= 19
       0  39.206  37.598  40.026  39.993  40.748  51.247  41.175  59.646  36.778
  65.715  30.577  75.492  29.593  95.571  27.723 107.808  27.297 118.471  31.234
 121.818  34.416 128.543  36.122 145.833  37.861 159.416  37.664 165.125  37.959
 173.031  41.667 180.643  42.093 193.963   39.37 220.079  39.304
#Mann= 3 , 0 , 0
       0    .035       0       0    .035       0 220.079    .035       0
Bank Sta=0,220.079
XS Rating Curve= 0
Exp/Cntr=.3,.1

Type RM Length L Ch R = 1 ,651     ,64.501,64.501,64.501
XS GIS Cut Line= 2
      5309703.67     15925023.69      5309921.62     15925134.74
#Sta/Elev= 20
       0  39.633  53.675  40.682  64.698  40.518  65.682   41.01  72.999   40.42
  81.365  34.875   85.63  31.135  91.043  29.593 113.944   27.92 132.316  27.756
 142.224  32.119 144.652  35.171 155.151   36.45 170.636   37.73 184.514  37.959
 189.665  40.846 191.732  41.535  203.15  41.634 216.765  40.387 244.619  39.042
#Mann= 3 , 0 , 0
       0    .035       0       0    .035       0 244.619    .035       0
Bank Sta=0,244.619
XS Rating Curve= 0
Exp/Cntr=.3,.1

Type RM Length L Ch R = 1 ,650     ,80.774,80.774,80.774
XS GIS Cut Line= 2
      5309687.86     15925058.53      5309842.81     15925193.21
#Sta/Elev= 18
       0  40.289   42.29  42.192  57.054  42.552  66.667  37.992  79.495  35.105
  81.923   31.43  85.335  29.626 107.054  28.084 127.756  28.215 131.529  31.299
 134.186  34.449 153.182  36.122 170.735  38.812 171.686  37.894  173.13  38.156
 177.657  40.945 182.087  41.634 205.315  42.126
#Mann= 3 , 0 , 0
       0    .035       0       0    .035       0 205.315    .035       0
Bank Sta=0,205.315
XS Rating Curve= 0
Exp/Cntr=.3,.1

Type RM Length L Ch R = 1 ,649     ,144.685,144.685,144.685
XS GIS Cut Line= 2
      5309665.55     15925065.58      5309734.97     15925267.13
#Sta/Elev= 18
       0  40.551  37.861  43.045    52.1  42.881  59.416  41.404  74.967  38.517
  88.911  35.991  94.291  31.988  99.836  29.462 115.354  27.986 137.795  29.298
  143.93  31.398 145.538  32.513 150.656  35.269 165.026  36.417 168.734  37.172
 171.982  40.617 183.169  42.028 213.156  40.551
#Mann= 3 , 0 , 0
       0    .035       0       0    .035       0 213.156    .035       0
Bank Sta=0,213.156
XS Rating Curve= 0
Exp/Cntr=.3,.1

Type RM Length L Ch R = 1 ,648     ,62.205,62.205,62.205
XS GIS Cut Line= 2
      5309561.58     15925048.46      5309565.35     15925265.22
#Sta/Elev= 19
       0    39.6  45.308   42.06  60.958  42.126  62.762  42.651  75.722  39.075
   83.99  37.795  92.848  36.417  99.442  33.038 100.886  31.496 107.513  28.839
 124.016  27.887 145.571  28.773 156.168  30.971 158.825  33.694 174.672  36.647
 182.185   40.65 193.373  40.912  194.98  39.993 216.798  39.272
#Mann= 3 , 0 , 0
       0    .035       0       0    .035       0 216.798    .035       0
Bank Sta=0,216.798
XS Rating Curve= 0
Exp/Cntr=.3,.1

Type RM Length L Ch R = 1 ,647     ,69.357,69.357,69.357
XS GIS Cut Line= 2
      5309493.11     15925050.43      5309500.82     15925271.42
#Sta/Elev= 18
       0  38.484  35.958  40.715  41.732   42.06  56.824  41.765  72.113   37.73
  84.547  36.778  89.534  33.727  91.109  31.824 102.526   28.51 119.619  27.822
 141.076  28.543  148.13  30.643 152.822  35.597 166.371  37.566  176.28  41.864
 191.667  41.929  193.57  39.534 221.129  39.862
#Mann= 3 , 0 , 0
       0    .035       0       0    .035       0 221.129    .035       0
Bank Sta=0,221.129
XS Rating Curve= 0
Exp/Cntr=.3,.1

Type RM Length L Ch R = 1 ,646     ,89.567,89.567,89.567
XS GIS Cut Line= 2
      5309412.47     15925047.51      5309440.75     15925277.85
#Sta/Elev= 17
       0  38.944  45.833  40.289  49.508  41.535  65.223  41.437  69.718  38.156
  88.451  36.417  95.079   33.99    97.9  31.496 109.744  28.182 131.004  27.756
 148.491  28.314 152.657  31.529 155.151  34.449 179.593  39.042 185.138  41.765
  200.82  41.306 232.087  39.961
#Mann= 3 , 0 , 0
       0    .035       0       0    .035       0 232.087    .035       0
Bank Sta=0,232.087
XS Rating Curve= 0
Exp/Cntr=.3,.1

Type RM Length L Ch R = 1 ,645     ,106.66,106.66,106.66
XS GIS Cut Line= 2
      5309313.02     15925071.78      5309354.43     15925251.18
#Sta/Elev= 14
       0  39.567   43.57  37.992  50.164  41.929  61.286  41.667   71.85  36.811
  84.022    35.4  89.272  30.118  96.358  27.887 120.833  27.723 133.629  28.084
 138.747  31.266  142.06  34.121 179.003  39.304 184.121  41.437
#Mann= 3 , 0 , 0
       0    .035       0       0    .035       0 184.121    .035       0
Bank Sta=0,184.121
XS Rating Curve= 0
Exp/Cntr=.3,.1

Type RM Length L Ch R = 1 ,644     ,89.567,89.567,89.567
XS GIS Cut Line= 2
      5309199.77     15925111.68      5309271.36     15925308.33
#Sta/Elev= 20
       0  38.484   34.35  37.959  40.354  40.978  52.329  41.207  55.052  39.764
  57.349  39.436   59.81   37.27  71.325  35.499  75.722   31.07  86.483  29.724
 109.252  27.461 120.243  29.199 127.231  31.135  132.71  35.105 171.654  39.993
 177.067  42.421 184.974   42.52 189.698  40.223 192.881  40.059 209.285  40.059
#Mann= 3 , 0 , 0
       0    .035       0       0    .035       0 209.285    .035       0
Bank Sta=0,209.285
XS Rating Curve= 0
Exp/Cntr=.3,.1

Type RM Length L Ch R = 1 ,643     ,61.713,61.713,61.713
XS GIS Cut Line= 2
      5309124.93     15925149.25       5309173.2     15925317.55
#Sta/Elev= 17
       0  41.207  19.718  41.798  22.703  42.946  32.349  42.979  41.798  37.992
  49.475  37.861  60.761   31.07  68.734  30.938  89.698  27.559 106.496   30.02
 112.664  30.938 117.848  35.794 128.379  37.533 152.592  40.026  161.22  44.226
 168.373  44.193 175.098  40.486
#Mann= 3 , 0 , 0
       0    .035       0       0    .035       0 175.098    .035       0
Bank Sta=0,175.098
XS Rating Curve= 0
Exp/Cntr=.3,.1

Type RM Length L Ch R = 1 ,642     ,22.014,22.014,22.014
XS GIS Cut Line= 2
      5309074.67     15925184.15       5309114.7     15925357.55
#Sta/Elev= 15
       0   45.44  16.404  45.472  26.706  36.319  37.238  34.777  40.715  31.398
  50.558  31.398  70.702  27.428  94.029  30.381 100.295  31.365 108.366  35.531
 119.948    37.5 125.459  39.206 134.121  45.407 143.504  45.866 177.953  44.488
#Mann= 3 , 0 , 0
       0    .035       0       0    .035       0 177.953    .035       0
Bank Sta=0,177.953
XS Rating Curve= 0
Exp/Cntr=.3,.1

Type RM Length L Ch R = 1 ,498.8   ,16.404,16.404,16.404
#Sta/Elev= 15
       0  46.522  72.375  46.752  85.728  36.155  94.783  35.269 101.214  31.594
 106.463  30.774 115.912  30.545 132.808  30.184 141.929  29.954 148.524   29.79
 154.757   31.43 164.665   35.63 172.867  36.417 187.434  46.752 221.883  45.374
#Mann= 3 , 0 , 0
       0    .035       0       0    .035       0 221.883    .035       0
Bank Sta=0,221.883
XS Rating Curve= 0
Exp/Cntr=.3,.1

Type RM Length L Ch R = 3 ,498.7   ,,,
BEGIN DESCRIPTION:
Ponte Salissimo
END DESCRIPTION:
Bridge Culvert--1,0,-1,-1, 0
Deck Dist Width WeirC Skew NumUp NumDn MinLoCord MaxHiCord MaxSubmerge Is_Ogee
1.64,13.123,2.61,0, 14, 14, , , .95, 0, 0,0,,
  72.375  85.728  85.728 111.024 111.024 115.584 115.584 141.929 141.929 146.916
 146.916 172.867 172.867 187.434
  46.752  46.752  46.752  46.752  46.752  46.752  46.752  46.752  46.752  46.752
  46.752  46.752  46.752  46.752
  46.752  36.155  43.176  43.209  30.676  30.545  43.209  43.209  29.954  29.823
  43.209  43.012  36.417  46.752
  72.375  85.728  85.728 111.024 111.024 115.584 115.584 141.929 141.929 146.916
 146.916 172.867 172.867 187.434
  46.752  46.752  46.752  46.752  46.752  46.752  46.752  46.752  46.752  46.752
  46.752  46.752  46.752  46.752
  46.752  36.155  43.176  43.209  30.676  30.545  43.209  43.209  29.954  29.823
  43.209  43.012  36.417  46.752
BR Coef=-1 , 0 , 0 ,1.25, 0 ,,,.8,-1,2,0,
WSPro=,,,, 1 ,,,, 0 ,,,, 0 ,,,,-1 ,-1 ,-1 , 0 , 0 , 0 , 0 , 0
BC Design=,, 0 ,, 0 ,,,,,,
BC HTab Sub Flow Pts= 40

Type RM Length L Ch R = 1 ,498.5   ,5.085,5.085,5.085
#Sta/Elev= 15
       0  46.522  72.375  46.752  85.728  36.155  94.783  35.269 101.214  31.594
 106.463  30.774 115.912  30.545 132.808  30.184 141.929  29.954 148.524   29.79
 154.757   31.43 164.665   35.63 172.867  36.417 187.434  46.752 221.883  45.374
#Mann= 3 , 0 , 0
       0    .035       0       0    .035       0 221.883    .035       0
Bank Sta=0,221.883
XS Rating Curve= 0
Exp/Cntr=.3,.1

Type RM Length L Ch R = 1 ,498     ,15.781,15.781,15.781
XS GIS Cut Line= 3
      5309047.47     15925174.15      5309086.65     15925331.04
      5309086.65     15925331.04
#Sta/Elev= 21
       0  46.575  22.762   46.45  32.031  46.004  46.276  35.207  57.054  35.049
  60.509  32.785  63.901  31.499   72.69  30.679  77.369  30.315  85.226   30.01
  88.343  29.948  93.018  29.774 100.233  29.846 103.993  30.423 108.921  30.781
 117.799  31.342 122.352  33.169 135.075  35.925 142.238  38.061 149.928  45.259
  163.13  45.052
#Mann= 3 , 0 , 0
       0    .035       0       0    .035       0  163.13    .035       0
Bank Sta=0,163.13
XS Rating Curve= 0
Exp/Cntr=.3,.1

Type RM Length L Ch R = 6 ,497.55  ,,,
Lateral Weir Pos= 3
Lateral Weir End=                ,                ,        ,c05
Lateral Weir Distance=3.281
Lateral Weir WD=9.843
Lateral Weir Coef=3.01
Lateral Weir Is Ogee= 0
Lateral Weir WSCriteria=-1
Lateral Weir SE= 6
       0   49.21    3.28   49.21    3.28   41.31  167.25   41.31  167.25   49.21
   171.5   49.21

Type RM Length L Ch R = 1 ,497     ,43.668,43.668,43.668
XS GIS Cut Line= 2
       5309037.4     15925176.64      5309073.06      15925337.3
#Sta/Elev= 23
       0  46.673  13.392  45.843  14.872  39.718   25.23  38.258  25.367  45.991
  31.896  45.978  32.418  36.919  35.377  36.736  38.678  34.836  59.501  35.118
  62.779  33.868  67.569  31.155   72.68  30.554  83.881  28.504  92.129  28.822
  96.739  29.436 112.726  30.541 117.018  32.566 128.136  34.918 141.539  37.077
 150.233  44.413 159.862  44.436 165.482  42.146
#Mann= 3 , 0 , 0
       0    .035       0       0    .035       0 165.482    .035       0
Bank Sta=0,165.482
XS Rating Curve= 0
Exp/Cntr=.3,.1

Type RM Length L Ch R = 1 ,496.5   ,85.86,85.86,85.86
XS GIS Cut Line= 2
      5308987.01     15925169.23      5309034.97     15925353.48
#Sta/Elev= 27
       0  41.785   32.92  41.017  35.502  40.528  41.719  43.527  46.365  43.668
  49.623   42.94  58.671  37.323  73.389  35.719  81.739  33.753  84.852  31.332
  87.972  29.475  90.108   28.78   96.44  27.736  103.34   26.47 113.166  26.224
 121.047  27.024 128.668  27.556 134.108  29.455 135.974  30.318 136.631   32.09
 142.326  32.808  144.82  34.403 151.985  35.558 165.194  36.168   172.5  41.864
 184.049  41.909 190.912  40.039
#Mann= 3 , 0 , 0
       0    .035       0       0    .035       0 190.912    .035       0
Bank Sta=0,190.912
XS Rating Curve= 0
Exp/Cntr=.3,.1

Type RM Length L Ch R = 1 ,496     ,161.155,161.155,161.155
XS GIS Cut Line= 2
      5308908.37      15925226.8      5308955.54     15925384.28
#Sta/Elev= 21
       0  37.526   8.983  37.612  15.479  40.722  19.098  40.545  25.062  34.895
  29.377  35.013  50.226  32.867  55.705   31.27  62.116  30.197  74.032  28.045
  82.982  27.559  90.951  27.546 100.541  30.774  103.13  33.885 118.202  35.456
 135.899  35.883 145.919  40.659 155.554  40.896 160.768  36.952 162.451  37.221
 164.793   39.82
#Mann= 3 , 0 , 0
       0    .035       0       0    .035       0 164.793    .035       0
Bank Sta=0,164.793
XS Rating Curve= 0
Exp/Cntr=.3,.1

Type RM Length L Ch R = 1 ,495     ,25.394,25.394,25.394
XS GIS Cut Line= 3
      5308740.12     15925246.72      5308824.28     15925494.91
      5308824.28     15925494.91
#Sta/Elev= 24
       0  40.748  27.684  40.279  39.154  39.049  45.627  37.871  54.567  36.188
  63.766  36.112  84.613  33.944  94.186  31.296  100.18  28.514 108.576   26.85
 113.822  26.854  125.22  30.161 130.682  30.846 140.469  32.326 142.133  33.615
 151.811  35.377 172.356  36.598 181.493  40.673 189.206   40.84 196.555  36.434
 198.268  36.168 199.918   37.74 237.208  38.642 262.871   38.74
#Mann= 3 , 0 , 0
       0    .035       0       0    .035       0 262.871    .035       0
Bank Sta=0,262.871
XS Rating Curve= 0
Exp/Cntr=.3,.1

Type RM Length L Ch R = 1 ,494     ,92.881,92.881,92.881
XS GIS Cut Line= 2
      5308715.26     15925266.17      5308785.76     15925440.45
#Sta/Elev= 22
       0  41.132   29.56  41.827  40.607  42.523  46.168  42.146  55.328  36.995
  66.631  35.702  78.087  33.842  84.724   30.86  89.278  31.204  96.237  31.155
 103.041  31.168 110.499  31.148  115.63  31.224  125.82   30.43 130.715  31.237
 154.229  30.456 171.791  31.824 172.372  40.922 176.847  41.283 180.358  42.382
  180.86  32.461 188.839  32.169
#Mann= 3 , 0 , 0
       0    .035       0       0    .035       0 180.358    .035       0
Bank Sta=0,180.358
XS Rating Curve= 0
Exp/Cntr=.3,.1

Type RM Length L Ch R = 6 ,493.55  ,,,
Lateral Weir Pos= 0
Lateral Weir End=                ,                ,        ,c06
Lateral Weir Distance=3.281
Lateral Weir WD=9.843
Lateral Weir Coef=3.01
Lateral Weir Is Ogee= 0
Lateral Weir WSCriteria=-1
Lateral Weir SE= 6
       0   49.21    3.28   49.21    3.28   41.31     330   41.31     330   49.21
  333.28   49.21

Type RM Length L Ch R = 1 ,493     ,229.79,229.79,229.79
XS GIS Cut Line= 2
      5308625.92     15925284.38      5308709.42     15925503.02
#Sta/Elev= 25
       0  39.147   25.41   39.82  47.382  36.043  51.532  35.443  52.385  42.769
  58.885  42.572  61.345  34.951  70.879  34.186   83.73   33.72  92.497  33.983
  99.439   32.68 102.812  29.354 107.552  30.784 114.154  29.439 122.913  27.149
 129.518  29.964 138.028   30.24 142.349  30.919 154.291  33.599 175.361  36.696
   187.1  41.985 191.033  41.969 199.049  38.783 213.727  39.432 234.895  39.147
#Mann= 3 , 0 , 0
       0    .035       0       0    .035       0 234.895    .035       0
Bank Sta=0,234.895
XS Rating Curve= 0
Exp/Cntr=.3,.1

Type RM Length L Ch R = 1 ,492     ,138.091,138.091,138.091
XS GIS Cut Line= 2
       5308414.4     15925350.26      5308491.63       15925596.
#Sta/Elev= 29
       0  39.649  34.465  40.167   56.03  36.503  57.503  40.584  64.957  41.089
  68.481  40.108  69.367  39.865  71.089  35.778  77.756  35.778  94.347  34.554
 109.583  33.547 113.363  32.697 116.568  30.715 120.236  30.883 127.451  30.814
 135.003  30.121 143.346  28.648  150.01  28.776 156.276   29.16 160.144  29.892
 161.063  31.896  167.11  32.969 174.455  36.765 182.894  37.694 190.738  41.099
 199.567  41.585   207.1  39.446 226.325  39.016 258.917  38.953
#Mann= 3 , 0 , 0
       0    .035       0  64.957    .035       0 199.567    .035       0
Bank Sta=64.957,199.567
XS Rating Curve= 0
Exp/Cntr=.3,.1

Type RM Length L Ch R = 1 ,491     ,174.442,174.442,174.442
XS GIS Cut Line= 2
      5308300.98     15925435.96      5308361.42     15925645.41
#Sta/Elev= 25
       0  35.919   2.241   39.79   5.322  41.175   8.671  41.342  11.785  40.308
  15.052  38.773  16.398  35.646  45.584  33.907  51.998  33.583    59.4  31.444
  69.386  30.932  75.955  29.606  81.319   27.47  87.073  27.113  94.304  26.512
 101.145  27.976 107.802  30.988 112.464  34.357 121.086  34.865 127.743  38.196
 137.014   41.68 144.839  41.499 151.785  39.173 181.316  38.173 218.763   38.51
#Mann= 3 , 0 , 0
       0    .035       0       0    .035       0 218.763    .035       0
Bank Sta=0,218.763
XS Rating Curve= 0
Exp/Cntr=.3,.1

Type RM Length L Ch R = 1 ,490     ,160.072,160.072,160.072
XS GIS Cut Line= 2
      5308119.69     15925407.97      5308195.34     15925690.26
#Sta/Elev= 23
       0  39.459  30.328  39.747  59.918  40.121  64.094  41.719  69.606  42.096
  74.954  40.988  82.287  36.988 103.268    34.6 120.856  34.042 127.014  32.464
 130.981  30.768 136.749  30.469  143.77  29.114  145.86  28.143 157.257  27.129
 175.325  31.056  180.42  34.321 191.864  36.056 203.888  41.709 211.398  42.146
 237.444  40.384 267.241  40.341 293.274   40.39
#Mann= 3 , 0 , 0
       0    .035       0       0    .035       0 293.274    .035       0
Bank Sta=0,293.274
XS Rating Curve= 0
Exp/Cntr=.3,.1

Type RM Length L Ch R = 1 ,489     ,147.178,147.178,147.178
XS GIS Cut Line= 3
      5307956.92     15925490.52      5308071.62     15925722.11
      5308071.62     15925722.11
#Sta/Elev= 25
       0  38.967  25.581  39.281  39.157  39.521  42.959  40.226  50.174  40.007
  54.409  39.219  59.826  36.677  70.315  34.895  85.449  33.665  89.491  31.417
  94.203  29.154  99.373  28.133 107.789  27.119 116.033  27.812 126.001  30.732
 130.144  31.066 136.591  30.974 145.876  34.183  166.27  36.394 170.522  36.952
 182.096  41.627 193.714  42.077 196.673  41.296 228.363  40.177 259.921  40.082
#Mann= 3 , 0 , 0
       0    .035       0       0    .035       0 259.921    .035       0
Bank Sta=0,259.921
XS Rating Curve= 0
Exp/Cntr=.3,.1

Type RM Length L Ch R = 1 ,488     ,171.129,171.129,171.129
XS GIS Cut Line= 2
      5307819.59     15925616.67      5307988.94     15925784.22
#Sta/Elev= 26
       0  40.758  13.632  40.141  20.846   37.91  36.319  37.677  38.071  42.703
  43.816  42.402  45.082  35.692  54.951  33.632  62.411  31.801  62.874  30.843
   67.92  29.938  74.803  27.779  83.727  26.778  89.344  30.394  93.415   31.03
  97.759   31.69 112.254   32.09  124.14   32.06 137.313  36.893 155.486  38.556
  167.73  40.318 172.772   42.11 178.455  42.297   179.6  41.621 207.769  40.131
 239.623  39.777
#Mann= 3 , 0 , 0
       0    .035       0       0    .035       0 239.623    .035       0
Bank Sta=0,239.623
XS Rating Curve= 0
Exp/Cntr=.3,.1

Type RM Length L Ch R = 1 ,487     ,154.396,154.396,154.396
XS GIS Cut Line= 2
      5307711.75     15925749.21      5307877.36       15925904.
#Sta/Elev= 21
       0   41.27  23.323  41.145  27.215  41.115  30.338  39.944  35.617  36.358
  42.736  35.138  45.512  34.242  46.365  30.823  51.818  28.753  59.754  28.297
  67.772  27.123  74.386  29.921  83.317  30.568 106.027  32.336 117.133  35.581
  143.11  37.411 151.791  41.726 164.501  41.558 170.381  39.009 200.463  38.547
 227.047  38.661
#Mann= 3 , 0 , 0
       0    .035       0       0    .035       0 227.047    .035       0
Bank Sta=0,227.047
XS Rating Curve= 0
Exp/Cntr=.3,.1

Type RM Length L Ch R = 6 ,486.55  ,,,
Lateral Weir Pos= 0
Lateral Weir End=                ,                ,        ,c04
Lateral Weir Distance=3.281
Lateral Weir WD=9.843
Lateral Weir Coef=3.01
Lateral Weir Is Ogee= 0
Lateral Weir WSCriteria=-1
Lateral Weir SE= 6
       0   49.21    3.28   49.21    3.28      40     320      40     320   49.21
  323.28   49.21

Type RM Length L Ch R = 1 ,486     ,262.73,262.73,262.73
XS GIS Cut Line= 3
        5307602.     15925873.85      5307790.29     15926016.47
      5307790.29     15926016.47
#Sta/Elev= 27
       0  39.203  14.993  38.888  16.795  37.277  18.225  37.336  19.741  38.478
  30.144  38.688  38.202  35.705  49.462  34.245  50.899  33.419  52.684  31.175
  58.711  27.119  65.299   24.82  70.016  25.469  79.101  27.762  84.783  30.407
  91.207  30.876  95.184   31.85 105.095  31.982 119.908  36.417 135.531  36.276
  148.99  38.022 156.535  42.139 167.523  42.254 174.281  40.292 177.228   38.77
 207.106  38.907 237.536  39.295
#Mann= 3 , 0 , 0
       0    .035       0       0    .035       0 237.536    .035       0
Bank Sta=0,237.536
XS Rating Curve= 0
Exp/Cntr=.3,.1

Type RM Length L Ch R = 1 ,485     ,176.969,176.969,176.969
XS GIS Cut Line= 3
      5307492.03      15926131.1      5307670.28     15926203.51
      5307670.28     15926203.51
#Sta/Elev= 21
       0  40.469   26.44  40.896  32.408  40.394  36.348  36.421  46.037  35.269
  51.854  32.205  52.972   30.81  58.251  28.422  66.562   27.74  76.637  28.399
  86.194  30.384  97.625  30.354 103.051  30.046 112.497   30.39 128.622  30.518
 139.573  29.934 152.172  30.459 152.769  42.323 164.298  42.172  177.06  31.975
 192.927  31.739
#Mann= 3 , 0 , 0
       0    .035       0       0    .035       0 192.927    .035       0
Bank Sta=0,192.927
XS Rating Curve= 0
Exp/Cntr=.3,.1

Type RM Length L Ch R = 6 ,484.55  ,,,
Lateral Weir Pos= 3
Lateral Weir End=                ,                ,        ,c05
Lateral Weir Distance=3.281
Lateral Weir WD=9.843
Lateral Weir Coef=3.01
Lateral Weir Is Ogee= 0
Lateral Weir WSCriteria=-1
Lateral Weir SE= 6
       0   49.21    3.28   49.21    3.28   38.69  495.08   38.69  495.68   49.21
     499   49.21

Type RM Length L Ch R = 1 ,484     ,177.001,177.001,177.001
XS GIS Cut Line= 3
       5307408.6     15926253.08      5307578.58     15926391.21
      5307578.58     15926391.21
#Sta/Elev= 23
       0  40.617  14.495  40.778  29.127  40.915  35.502  40.604  39.692  40.262
  44.252  35.627  54.941  34.331   65.61  34.865  72.169  34.442  80.479  31.631
  81.453  30.666  86.014  30.069  90.269  28.412  96.752  26.112  107.74  26.788
 116.732   29.59 121.309  31.066 135.384  34.836 148.409  34.944 161.411  35.407
 166.693  36.667 194.409   38.12 219.268  38.996
#Mann= 3 , 0 , 0
       0    .035       0       0    .035       0 219.268    .035       0
Bank Sta=0,219.268
XS Rating Curve= 0
Exp/Cntr=.3,.1

Type RM Length L Ch R = 1 ,483     ,159.252,159.252,159.252
XS GIS Cut Line= 3
      5307294.09     15926340.68      5307420.47     15926534.02
      5307420.47     15926534.02
#Sta/Elev= 20
       0  40.794  21.732  41.047  40.276  40.538  49.685  34.455  58.996  33.776
   69.58  34.587  76.565   33.77  85.837  31.939  87.923  30.843  92.454  30.417
 100.404   27.07 107.467  26.447  114.15  26.112 119.491  27.434 124.665   30.24
 133.645   35.02 166.404  35.095 174.757  39.108 204.419  40.148 231.309  39.793
#Mann= 3 , 0 , 0
       0    .035       0       0    .035       0 204.419    .035       0
Bank Sta=0,204.419
XS Rating Curve= 0
Exp/Cntr=.3,.1

Type RM Length L Ch R = 1 ,482     ,202.953,202.953,202.953
XS GIS Cut Line= 2
       5307185.7     15926429.72       5307258.6     15926646.69
#Sta/Elev= 23
       0  39.984  12.277  39.993  20.354  34.783  31.142  33.576  38.665  33.182
  48.494  33.451  50.712  31.516  56.319  30.489  62.192  29.091  67.274  28.402
  76.352  28.727  83.573  30.056  88.688  30.719  95.335   31.22  98.537  32.001
 111.138  34.052 121.716   35.21  142.68  36.358 151.785  41.135 153.947  40.922
 155.922  39.678 205.633  39.629 229.282  39.564
#Mann= 3 , 0 , 0
       0    .035       0       0    .035       0 229.282    .035       0
Bank Sta=0,229.282
XS Rating Curve= 0
Exp/Cntr=.3,.1

Type RM Length L Ch R = 1 ,481     ,264.469,264.469,264.469
XS GIS Cut Line= 2
      5306991.31     15926446.26      5307037.66     15926688.06
#Sta/Elev= 22
       0  39.839  22.904  40.197  33.415  39.154  41.519  36.696  50.748  34.652
  72.818  33.678  84.357  33.737  89.603  31.476  96.152  30.056 105.682    28.1
  112.53  26.411 118.186  26.424 128.169  28.675 132.871  30.646 133.766  32.451
 141.952  34.495 155.302  35.646 157.201  36.608  178.36  39.554  181.65  39.114
 215.459  38.894 246.617  38.783
#Mann= 3 , 0 , 0
       0    .035       0       0    .035       0 246.617    .035       0
Bank Sta=0,246.617
XS Rating Curve= 0
Exp/Cntr=.3,.1

Type RM Length L Ch R = 1 ,480     ,145.571,145.571,145.571
XS GIS Cut Line= 3
      5306786.42      15926454.4      5306744.69     15926623.92
      5306744.69     15926623.92
#Sta/Elev= 22
       0  40.758  32.001  41.027  34.491  40.043  42.602   34.97  55.932  35.371
  66.634  35.696  73.816  34.357  82.175  33.625  88.921   31.07  98.248  30.774
 105.003   30.23 110.299  28.461 116.716  28.953 123.596  28.904 132.677  30.039
 137.405  30.135 148.812  30.692  155.83   30.19 156.657  42.828 162.133   42.72
 162.848   32.06 175.262  32.267
#Mann= 3 , 0 , 0
       0    .035       0       0    .035       0 175.262    .035       0
Bank Sta=0,175.262
XS Rating Curve= 0
Exp/Cntr=.3,.1

Type RM Length L Ch R = 6 ,479.55  ,,,
Lateral Weir Pos= 0
Lateral Weir End=                ,                ,        ,c04
Lateral Weir Distance=3.281
Lateral Weir WD=9.843
Lateral Weir Coef=3.01
Lateral Weir Is Ogee= 0
Lateral Weir WSCriteria=-1
Lateral Weir SE= 6
       0   49.21    3.28   49.21    3.28   39.67  167.32   39.67  167.32   49.21
   170.6   49.21

Type RM Length L Ch R = 1 ,479     ,171.654,171.654,171.654
XS GIS Cut Line= 2
      5306655.54      15926404.3      5306593.96     15926634.15
#Sta/Elev= 21
       0  43.389  44.209  42.703  52.247  37.562  63.747  36.998  78.406  36.998
  90.499  37.333  94.885   36.47  98.907  34.032  104.99  31.132  111.01  29.016
 117.972  27.441 126.683  27.438 136.545  28.796 140.751  30.069 144.121   34.37
  149.39  35.594 164.072  41.916 174.514  41.916 179.551  39.692  217.68  39.583
 238.468  39.708
#Mann= 3 , 0 , 0
       0    .035       0       0    .035       0 238.468    .035       0
Bank Sta=0,238.468
XS Rating Curve= 0
Exp/Cntr=.3,.1

Type RM Length L Ch R = 1 ,478     ,150.722,150.722,150.722
XS GIS Cut Line= 3
      5306487.04     15926364.63      5306420.87     15926573.85
      5306420.87     15926573.85
#Sta/Elev= 21
       0  39.596  28.376  39.846  41.535  33.645  56.775  33.776   76.66  34.905
  80.203  33.855  84.173  30.505  87.982  30.443  96.424  28.084 104.639  27.379
 110.755  26.834 116.588  27.379 123.176  29.524 126.903  30.587 132.306  34.245
 139.537  35.715 152.451  41.542 160.748  41.883 168.258  39.557 192.894  39.469
 220.016  39.413
#Mann= 3 , 0 , 0
       0    .035       0       0    .035       0 220.016    .035       0
Bank Sta=0,220.016
XS Rating Curve= 0
Exp/Cntr=.3,.1

Type RM Length L Ch R = 1 ,477     ,89.108,89.108,89.108
XS GIS Cut Line= 3
      5306343.96     15926322.44      5306294.82     15926490.35
      5306294.82     15926490.35
#Sta/Elev= 20
       0  41.161  20.489  41.883   24.97  41.463  41.444  33.593  55.482  34.232
  72.277  34.216  80.554  30.564  84.905  29.265  92.484  27.674  101.27  27.152
 110.285  27.986 116.132  27.825 124.974  29.774 128.589   32.69 140.751  33.563
 151.299  33.107 152.133  42.927 160.056  42.733 160.584   33.95 175.341  36.007
#Mann= 3 , 0 , 0
       0    .035       0       0    .035       0 175.341    .035       0
Bank Sta=0,175.341
XS Rating Curve= 0
Exp/Cntr=.3,.1

Type RM Length L Ch R = 1 ,476     ,165.19,165.19,165.19
XS GIS Cut Line= 3
      5306253.58      15926314.6      5306195.37     15926504.99
      5306195.37     15926504.99
#Sta/Elev= 21
       0  42.267   5.997  42.687   6.404  31.955  20.853  32.024  36.522  31.617
   44.36  32.339  49.393  32.881  52.188  31.355  58.045  30.784  65.059  28.438
  73.435  27.064  82.897  27.638  93.091  27.762 100.121  30.623 104.524   31.02
 115.725  37.051 126.696  38.757  130.23  40.784 143.786  40.571 174.452  39.196
 200.138  38.796
#Mann= 3 , 0 , 0
       0    .035       0       0    .035       0 200.138    .035       0
Bank Sta=0,200.138
XS Rating Curve= 0
Exp/Cntr=.3,.1

Type RM Length L Ch R = 1 ,475     ,218.766,218.766,218.766
XS GIS Cut Line= 3
      5306111.55     15926225.95      5306032.02     15926463.91
      5306032.02     15926463.91
#Sta/Elev= 25
       0  44.446  28.556  44.872  33.169  44.278  38.025   42.72  48.871  42.352
  59.469  36.919  68.809   35.85  78.658  33.921  85.942  31.969  88.727  31.165
  94.055   30.43 102.024  27.703 110.331  26.598 118.694  27.628 127.697  27.687
 133.271  30.338 137.907  30.843 144.574  33.757 152.733  37.096 169.888   38.74
 176.617  42.021 186.463  41.637 190.669  39.308 219.603  39.242 251.293  39.114
#Mann= 3 , 0 , 0
       0    .035       0       0    .035       0 251.293    .035       0
Bank Sta=0,251.293
XS Rating Curve= 0
Exp/Cntr=.3,.1

Type RM Length L Ch R = 1 ,474     ,169.291,169.291,169.291
XS GIS Cut Line= 2
      5305846.16     15926211.71      5305870.05     15926404.27
#Sta/Elev= 21
       0  40.066  27.178  41.427  34.409  40.951  40.302  40.597  56.631   35.44
  65.814  32.464  67.159  31.079   71.49  28.714  78.816  27.215   86.47  25.669
  96.411  27.464 103.553   29.39 113.963  30.449 120.568  30.919 130.056  33.018
 155.725  33.586 168.671   34.57 169.219  42.172  175.03  41.926 175.568  36.089
 194.836  38.327
#Mann= 3 , 0 , 0
       0    .035       0       0    .035       0 194.836    .035       0
Bank Sta=0,194.836
XS Rating Curve= 0
Exp/Cntr=.3,.1

Type RM Length L Ch R = 1 ,473.5   ,18.176,18.176,18.176
XS GIS Cut Line= 2
      5305669.98     15926267.65      5305729.23     15926456.73
#Sta/Elev= 23
       0  41.273   3.412  42.585  25.525  41.667  26.772  40.879  34.613  35.958
  43.307   34.81  51.837  31.135  58.825  29.954  62.631  28.773  67.093  27.789
  71.949  26.837  76.181  27.264  78.871  27.756  88.058  30.348   92.06  30.971
  97.211  30.807 101.214  31.037  105.61  31.726 123.524  39.993 141.306  40.978
 141.568   41.01 173.294  40.551 198.655  40.026
#Mann= 3 , 0 , 0
       0    .035       0  26.772    .035       0 141.306    .035       0
Bank Sta=26.772,141.306
XS Rating Curve= 0
Exp/Cntr=.3,.1

Type RM Length L Ch R = 1 ,473     ,26.739,26.739,26.739
XS GIS Cut Line= 2
      5305648.79     15926264.44      5305704.63     15926430.28
#Sta/Elev= 18
       0  44.291  16.207  44.751   41.01  45.571  41.109  45.472  54.364  35.039
  61.811  32.743  63.583  30.971  69.554  31.037   76.05  31.004  81.004  31.004
  91.437  31.004 107.119  30.381 112.664  31.824 122.507  35.597 135.138  45.308
 135.269   45.44 157.087  45.013 175.755  44.193
#Mann= 3 , 0 , 0
       0    .035       0  41.109    .035       0 135.138    .035       0
Bank Sta=41.109,135.138
XS Rating Curve= 0
Exp/Cntr=.3,.1

Type RM Length L Ch R = 1 ,472.9   ,32.808,32.808,32.808
XS GIS Cut Line= 2
      5305615.49      15926227.4       5305706.5     15926481.76
#Sta/Elev= 18
       0  44.816  42.028  46.293  52.165  45.669  64.993  35.958   76.05  32.382
  77.362  31.004  82.743  30.446  94.226  29.101 102.067  28.773 114.797  30.413
 118.602  30.873  126.28  34.285 132.513  36.909  144.39  45.308 145.276  45.965
 164.567  45.604 189.698   44.39 208.071   43.34
#Mann= 3 , 0 , 0
       0    .035       0       0    .035       0 208.071    .035       0
Bank Sta=0,208.071
XS Rating Curve= 0
Exp/Cntr=.3,.1

Type RM Length L Ch R = 3 ,472.8   ,,,
BEGIN DESCRIPTION:
ponte di meati
END DESCRIPTION:
Bridge Culvert--1,0,-1,-1, 0
Deck Dist Width WeirC Skew NumUp NumDn MinLoCord MaxHiCord MaxSubmerge Is_Ogee
1.64,29.528,2.61,0, 11, 11, , , .95, 0, 0,0,,
       0  42.028  52.133  64.895  64.895  82.021 132.382 132.382 164.337 189.501
 207.841
  47.113  47.113  47.113  47.113  47.113  47.113  47.113  47.113  47.113  47.113
  47.113
  41.306  41.306  41.306  35.958  41.306  41.306  41.306  36.909  41.306  41.306
  41.306
       0  42.028  52.133  64.895  64.895  82.021 132.382 132.382 164.337 189.501
 207.841
  47.113  47.113  47.113  47.113  47.113  47.113  47.113  47.113  47.113  47.113
  47.113
  41.306  41.306  41.306  35.958  41.306  41.306  41.306  36.909  41.306  41.306
  41.306
BR Coef=-1 , 0 , 0 ,1.25, 0 ,,,.8,-1,2,0,
WSPro=,,,, 1 ,,,, 0 ,,,, 0 ,,,,-1 ,-1 ,-1 , 0 , 0 , 0 , 0 , 0
BC Design=,, 0 ,, 0 ,,,,,,
BC HTab Sub Flow Pts= 40

Type RM Length L Ch R = 1 ,472.7   ,50.984,50.984,50.984
XS GIS Cut Line= 2
      5305615.49      15926227.4       5305706.5     15926481.76
#Sta/Elev= 18
       0  44.816  42.028  46.293  52.165  45.669  64.993  35.958   76.05  32.382
  77.362  31.004  82.743  30.446  94.226  29.101 102.067  28.773 114.797  30.413
 118.602  30.873  126.28  34.285 132.513  36.909  144.39  45.308 145.276  45.965
 164.567  45.604 189.698   44.39 208.071   43.34
#Mann= 3 , 0 , 0
       0    .035       0       0    .035       0 208.071    .035       0
Bank Sta=0,208.071
XS Rating Curve= 0
Exp/Cntr=.3,.1

Type RM Length L Ch R = 1 ,472     ,172.441,172.441,172.441
XS GIS Cut Line= 2
      5305550.98     15926224.02      5305615.78     15926497.93
#Sta/Elev= 20
       0  43.698  37.595  43.822  64.491   43.36  85.269  38.133 102.149  35.928
 115.738  32.018 116.506  31.647 124.911  30.446 137.621  27.805 144.511  29.131
 153.566  26.476 160.072   27.48 168.038  31.207 179.777  32.831 186.014  35.102
 205.719  34.895 225.525   34.97 241.906  39.068 257.746  40.341 281.693  40.745
#Mann= 3 , 0 , 0
       0    .035       0       0    .035       0 281.693    .035       0
Bank Sta=0,281.693
XS Rating Curve= 0
Exp/Cntr=.3,.1

Type RM Length L Ch R = 1 ,471     ,163.944,163.944,163.944
XS GIS Cut Line= 2
      5305388.19     15926311.09      5305461.15     15926532.61
#Sta/Elev= 21
       0  40.289  27.349  41.102  31.896  42.966  45.505  42.313  54.852  37.087
  67.972  35.541  74.685  31.532  81.112   30.44  91.906  27.493 102.441   25.85
 108.609  27.805 118.268  30.436 127.096  31.699 134.226  34.216  149.15  34.321
 169.829  34.275 190.968  35.046 203.212  35.581 213.773  35.745 220.686  35.633
 233.914  35.709
#Mann= 3 , 0 , 0
       0    .035       0       0    .035       0 233.914    .035       0
Bank Sta=0,233.914
XS Rating Curve= 0
Exp/Cntr=.3,.1

Type RM Length L Ch R = 1 ,470     ,123.458,123.458,123.458
XS GIS Cut Line= 2
      5305239.24      15926364.3      5305290.42     15926579.69
#Sta/Elev= 16
       0  33.875  22.385  33.599  41.411  33.255  59.393  31.309  65.673  29.455
  76.309  28.675  87.503  27.648  95.351  27.687 100.679  29.049 109.761  29.213
 116.867  33.868 136.952  33.652 158.852  33.789 171.673   34.57 189.938  39.895
 221.444  40.459
#Mann= 3 , 0 , 0
       0    .035       0       0    .035       0 221.444    .035       0
Bank Sta=0,221.444
XS Rating Curve= 0
Exp/Cntr=.3,.1

Type RM Length L Ch R = 6 ,469.55  ,,,
Lateral Weir Pos= 3
Lateral Weir End=                ,                ,        ,c01
Lateral Weir Distance=3.281
Lateral Weir WD=9.843
Lateral Weir Coef=3.01
Lateral Weir Is Ogee= 0
Lateral Weir WSCriteria=-1
Lateral Weir SE= 6
       0   49.21    3.28   49.21    3.28   37.73  331.37   37.73  331.37   49.21
  334.65   49.21

Type RM Length L Ch R = 1 ,469     ,225.23,225.23,225.23
XS GIS Cut Line= 2
      5305115.16     15926339.63      5305164.93     15926599.87
#Sta/Elev= 17
       0  38.658   52.73  38.258  77.854  37.274  91.644   35.62 118.235  34.065
 119.396  31.411 128.724  28.976 142.185   27.74 154.905  28.921 162.887  29.475
 169.895  30.646 173.629  33.871 190.679  33.842 203.816  33.645 215.105  35.787
 226.604  39.249 265.079  40.285
#Mann= 3 , 0 , 0
       0    .035       0       0    .035       0 265.079    .035       0
Bank Sta=0,265.079
XS Rating Curve= 0
Exp/Cntr=.3,.1

Type RM Length L Ch R = 6 ,468.55  ,,,
Lateral Weir Pos= 0
Lateral Weir End=                ,                ,        ,c02
Lateral Weir Distance=3.281
Lateral Weir WD=9.843
Lateral Weir Coef=3.01
Lateral Weir Is Ogee= 0
Lateral Weir WSCriteria=-1
Lateral Weir SE= 6
       0  49.213   3.281  49.213   3.281   41.01 987.533   41.01 987.533  49.213
 990.814  49.213

Type RM Length L Ch R = 1 ,468     ,87.828,87.828,87.828
XS GIS Cut Line= 3
      5304888.98     15926404.17      5304945.47      15926622.8
      5304945.47      15926622.8
#Sta/Elev= 22
       0  40.915  65.778   40.86  75.121   41.49  89.718  34.154 109.514  34.721
 112.995  33.346 114.334  30.584 120.272  27.946 130.148  28.691 137.533  27.841
 147.257  27.648 155.052  28.888 162.093  29.977 164.006  32.306 170.466  33.563
 181.132  34.101 188.136  34.721 196.591  36.883 202.986  42.073 206.932   42.09
 213.852  39.485 226.191  39.547
#Mann= 3 , 0 , 0
       0    .035       0       0    .035       0 226.191    .035       0
Bank Sta=0,226.191
XS Rating Curve= 0
Exp/Cntr=.3,.1

Type RM Length L Ch R = 1 ,467     ,83.53,83.53,83.53
XS GIS Cut Line= 3
      5304819.82     15926464.27      5304852.72     15926633.33
      5304852.72     15926633.33
#Sta/Elev= 19
       0  40.121  19.974  36.991  40.696  35.095  70.748  34.495  75.705  32.467
   77.06  30.919  81.755   30.42  89.649  27.224  96.102  28.865 102.812  27.349
 109.252  27.162 115.922  27.703 121.936  29.764 126.053  32.795 138.468  34.101
 151.975  35.771 163.625  42.762 168.209  42.467  172.51  41.083
#Mann= 3 , 0 , 0
       0    .035       0       0    .035       0  172.51    .035       0
Bank Sta=0,172.51
XS Rating Curve= 0
Exp/Cntr=.3,.1

Type RM Length L Ch R = 1 ,466     ,134.875,134.875,134.875
XS GIS Cut Line= 2
      5304737.83     15926472.28      5304795.77     15926720.34
#Sta/Elev= 18
       0   34.77  47.572  33.694   56.86  33.071  88.087  31.056  96.788  29.396
 103.002   26.85 109.665  26.499 116.198   26.66  122.73  26.854 128.599  29.606
 134.865  30.318 139.925  32.792 153.396  33.491 162.871  33.802 178.189  42.103
 186.076   42.49 192.861  39.816 255.902  39.843
#Mann= 3 , 0 , 0
       0    .035       0       0    .035       0 255.902    .035       0
Bank Sta=0,255.902
XS Rating Curve= 0
Exp/Cntr=.3,.1

Type RM Length L Ch R = 1 ,465     ,216.831,216.831,216.831
XS GIS Cut Line= 2
      5304594.72      15926531.5      5304671.13     15926729.07
#Sta/Elev= 20
       0  40.384  34.016  40.308  39.948  39.961  54.304  34.377  72.592  34.318
  74.948  33.622  76.007  31.122   82.28    27.5  89.734  26.112  96.542  26.099
 106.312  26.923 112.333  30.584 120.525  30.725 126.545  32.743 143.402  33.002
 155.052  33.583 166.562  33.451 174.865  34.892 190.384  35.453 212.136  35.653
#Mann= 3 , 0 , 0
       0    .035       0       0    .035       0 212.136    .035       0
Bank Sta=0,212.136
XS Rating Curve= 0
Exp/Cntr=.3,.1

Type RM Length L Ch R = 1 ,464     ,190.978,190.978,190.978
XS GIS Cut Line= 3
      5304372.74     15926566.11      5304488.16     15926855.64
      5304488.16     15926855.64
#Sta/Elev= 22
       0  39.452  56.736  40.492  84.423  40.804  88.648  40.361 105.246  34.672
 128.481  33.284 131.867  32.444 133.517   31.01 138.763  28.448 146.496  26.506
  153.31   26.45 159.688  26.565  166.45   26.68 170.899   28.72 177.792  30.476
 184.147  33.629 198.937  33.114 217.208  42.129  223.32  42.192 230.305  40.246
 242.831   40.22 311.778  39.967
#Mann= 3 , 0 , 0
       0    .035       0       0    .035       0 311.778    .035       0
Bank Sta=0,311.778
XS Rating Curve= 0
Exp/Cntr=.3,.1

Type RM Length L Ch R = 1 ,463     ,186.483,186.483,186.483
XS GIS Cut Line= 3
      5304196.23     15926644.78      5304288.35     15926877.82
      5304288.35     15926877.82
#Sta/Elev= 22
       0  40.367  57.428  41.053  80.443  40.492  98.028  33.868 109.587  33.422
 123.717  33.858 128.612  30.958 134.432  29.843 142.874  26.736 152.477  26.201
 159.176  26.001 167.139  27.251 172.631  28.967 176.102  32.021 187.585  33.219
 199.173  33.202 207.644  34.993 208.835  42.073 217.198  41.765 217.526  35.335
 234.032  36.785 251.089  37.346
#Mann= 3 , 0 , 0
       0    .035       0       0    .035       0 251.089    .035       0
Bank Sta=0,251.089
XS Rating Curve= 0
Exp/Cntr=.3,.1

Type RM Length L Ch R = 1 ,462     ,164.206,164.206,164.206
XS GIS Cut Line= 2
        5304025.     15926723.88      5304128.44     15926964.63
#Sta/Elev= 24
       0  39.442  55.266  39.941  61.965  43.087  66.001   42.71  70.482  41.434
  85.489  33.514 111.716  33.232 113.825  34.134 118.612  32.835 119.439  30.617
 125.699  28.865 133.783  27.441 143.261  25.505 149.846  25.971 156.526  27.211
 159.669  29.715  163.15  29.911 165.305  32.487 181.729  33.878  198.53  42.398
  204.35  42.159 211.604  40.161 231.509  39.803 262.238  39.921
#Mann= 3 , 0 , 0
       0    .035       0       0    .035       0 262.238    .035       0
Bank Sta=0,262.238
XS Rating Curve= 0
Exp/Cntr=.3,.1

Type RM Length L Ch R = 1 ,461     ,106.759,106.759,106.759
XS GIS Cut Line= 2
      5303893.57     15926821.19      5303982.84     15927045.87
#Sta/Elev= 23
       0  39.705  21.558  37.884  28.264  35.443  32.113  38.704  38.871   39.79
  41.401  34.777  49.055   33.32  78.563  32.421  80.394  30.607  87.093  28.002
  92.559  26.745 102.343  26.585 108.957  26.706 115.623  27.464  120.81  29.593
 124.787  30.171 127.657  31.932 150.023  33.602  164.81  42.349 168.307  42.405
 173.465  41.358 197.894  40.945 243.002  40.315
#Mann= 3 , 0 , 0
       0    .035       0       0    .035       0 243.002    .035       0
Bank Sta=0,243.002
XS Rating Curve= 0
Exp/Cntr=.3,.1

Type RM Length L Ch R = 1 ,460     ,215.814,215.814,215.814
XS GIS Cut Line= 3
      5303770.34     15926850.69       5303876.8     15927054.92
       5303876.8     15927054.92
#Sta/Elev= 21
       0   39.78  52.392  40.528  55.614  42.221   66.86  41.929  79.505  34.367
 100.591  33.691 103.743   31.27 110.984  28.215 118.156  26.801 125.016   26.44
 131.473  26.745 138.369  28.015 145.433  29.816 152.536  30.584 156.614  32.421
 179.229  33.094 193.734  35.089 194.475  42.543 200.312  42.461 200.502  36.283
 231.532  36.903
#Mann= 3 , 0 , 0
       0    .035       0       0    .035       0 231.532    .035       0
Bank Sta=0,231.532
XS Rating Curve= 0
Exp/Cntr=.3,.1

Type RM Length L Ch R = 6 ,459.55  ,,,
Lateral Weir Pos= 0
Lateral Weir End=                ,                ,        ,c02
Lateral Weir Distance=3.281
Lateral Weir WD=9.843
Lateral Weir Coef=3.01
Lateral Weir Is Ogee= 0
Lateral Weir WSCriteria=-1
Lateral Weir SE= 6
       0  49.213   3.281  49.213   3.281  42.323 167.323  42.323 167.323  49.213
 170.604  49.213

Type RM Length L Ch R = 1 ,459     ,132.874,132.874,132.874
XS GIS Cut Line= 2
      5303607.55     15926978.05      5303688.68     15927175.56
#Sta/Elev= 23
       0  39.974  11.667   36.22  18.763  34.715  20.308   40.43  20.866  34.783
  30.912  34.183   31.86  34.032  54.875  33.983  66.909  33.419  72.215  32.067
  72.953  30.771  79.196  29.869  87.851  27.474  94.505  25.997 100.978   27.07
 103.842  27.323 113.714  29.413 116.119  31.795 123.953  33.271 141.234  33.615
 156.909  41.798 177.753  42.703 215.935  42.484
#Mann= 3 , 0 , 0
       0    .035       0       0    .035       0 215.935    .035       0
Bank Sta=0,215.935
XS Rating Curve= 0
Exp/Cntr=.3,.1

Type RM Length L Ch R = 1 ,458     ,150.066,150.066,150.066
XS GIS Cut Line= 2
      5303493.31     15927073.49      5303597.18     15927255.18
#Sta/Elev= 16
       0  35.604   9.295  34.272  35.971  33.802  42.671  31.158  50.863  29.032
  61.755    26.9  71.808  27.454  79.108  28.179  84.741  28.727  88.133  29.498
  94.678  33.993 120.236  36.047 131.867  42.129 137.664   43.15 177.451   42.73
 209.633  42.779
#Mann= 3 , 0 , 0
       0    .035       0       0    .035       0 209.633    .035       0
Bank Sta=0,209.633
XS Rating Curve= 0
Exp/Cntr=.3,.1

Type RM Length L Ch R = 1 ,457     ,108.924,108.924,108.924
XS GIS Cut Line= 2
      5303325.66      15927097.9       5303451.8     15927284.28
#Sta/Elev= 21
       0  42.697  40.843  42.802  76.535  41.293  90.407  33.668 112.963  33.757
  115.18  31.562 120.981  27.365 128.816  25.974 135.381  25.387 141.729  25.256
 150.686  29.045 155.863  30.407 159.442    29.6 163.484  32.621 174.304  33.182
 195.886  33.468 200.479  35.246 201.132  42.969 207.228  42.779 207.766  37.323
 225.256  39.272
#Mann= 3 , 0 , 0
       0    .035       0       0    .035       0 225.256    .035       0
Bank Sta=0,225.256
XS Rating Curve= 0
Exp/Cntr=.3,.1

Type RM Length L Ch R = 1 ,456     ,137.73,137.73,137.73
XS GIS Cut Line= 3
      5303269.65     15927219.06        5303375.     15927382.81
        5303375.     15927382.81
#Sta/Elev= 18
       0  37.677  10.351  36.171  19.833  34.701  43.432  33.255  45.374  30.479
  51.923  28.937  59.462  26.713   66.03  26.204  76.033  26.312  83.891  27.274
  88.862   29.35  94.478  31.788 101.476  33.894 116.752   33.96 134.012  42.244
 145.108  43.422 177.717  43.533 197.047  43.392
#Mann= 3 , 0 , 0
       0    .035       0       0    .035       0 197.047    .035       0
Bank Sta=0,197.047
XS Rating Curve= 0
Exp/Cntr=.3,.1

Type RM Length L Ch R = 1 ,455     ,262.336,262.336,262.336
XS GIS Cut Line= 3
      5303150.98     15927298.62       5303289.8     15927460.37
       5303289.8     15927460.37
#Sta/Elev= 17
       0  34.715  11.083  34.108  20.741  32.152  28.822  32.041  45.154   32.29
  51.332  31.109   59.14  29.606  65.512  26.926  75.322  26.716  81.949  26.854
  90.456  28.691  95.282  29.619 100.479  33.543 127.103  34.285 142.651  42.749
 166.893  43.159 213.917  42.743
#Mann= 3 , 0 , 0
       0    .035       0       0    .035       0 213.917    .035       0
Bank Sta=0,213.917
XS Rating Curve= 0
Exp/Cntr=.3,.1

Type RM Length L Ch R = 1 ,454     ,198.72,198.72,198.72
XS GIS Cut Line= 2
      5302932.25     15927384.42      5303022.41     15927574.74
#Sta/Elev= 20
       0  46.722  50.482  47.224  57.434  43.035  71.837  42.615  82.028  36.135
 109.836  35.308 117.195  33.287 121.673  30.889 131.447  30.043 137.927  28.399
 144.551  26.788 151.325  26.696 157.966  25.961 165.879  28.205 170.643  30.036
 175.062  33.369 189.977  34.659 201.178  41.709 204.902  42.398 210.912  42.369
#Mann= 3 , 0 , 0
       0    .035       0       0    .035       0 210.912    .035       0
Bank Sta=0,210.912
XS Rating Curve= 0
Exp/Cntr=.3,.1

Type RM Length L Ch R = 6 ,453.55  ,,,
Lateral Weir Pos= 3
Lateral Weir End=                ,                ,        ,c01
Lateral Weir Distance=3.281
Lateral Weir WD=9.843
Lateral Weir Coef=3.01
Lateral Weir Is Ogee= 0
Lateral Weir WSCriteria=-1
Lateral Weir SE= 6
       0  49.213   3.281  49.213   3.281  41.667 331.365  41.667 331.365  49.213
 334.646  49.213

Type RM Length L Ch R = 1 ,453     ,159.908,159.908,159.908
XS GIS Cut Line= 2
      5302774.28     15927435.63      5302813.58     15927638.16
#Sta/Elev= 29
       0  43.041  10.666  40.758  14.022  40.387  23.832  44.774  32.579      50
  36.411  50.115  46.532  43.583  61.939  42.995  70.505  36.745  99.108  34.951
  112.48  31.309 123.117  30.741  130.64   27.74 136.995  25.709 143.707  25.459
 150.479  26.024 155.732  27.438 160.909  29.649 162.569   32.89 166.952  34.232
 182.077  35.541 190.919  40.965 194.685  42.339 198.842  43.028 204.928  45.797
 205.167  47.927 205.971   47.92 206.099  48.625 208.058  48.976
#Mann= 3 , 0 , 0
       0    .035       0       0    .035       0 208.058    .035       0
Bank Sta=0,208.058
XS Rating Curve= 0
Exp/Cntr=.3,.1

Type RM Length L Ch R = 1 ,452     ,7.251,7.251,7.251
XS GIS Cut Line= 2
      5302612.43     15927499.18      5302673.56       15927644.
#Sta/Elev= 22
       0  40.545   8.209  39.997  18.504  36.263  40.591  36.043  42.218  45.676
  42.904  45.699  43.219  43.458  48.038  43.396  48.694  45.709  49.465  45.735
  50.607  33.793  56.155  31.749  75.705  30.761  82.011  28.123  90.554  27.388
 100.374  28.474 107.014  28.379 116.188   30.44  119.61  30.554 122.146  32.785
 137.894   33.36  161.64  33.766
#Mann= 3 , 0 , 0
       0    .035       0       0    .035       0  161.64    .035       0
Bank Sta=0,161.64
XS Rating Curve= 0
Exp/Cntr=.3,.1

Type RM Length L Ch R = 1 ,451     ,15.748,15.748,15.748
XS GIS Cut Line= 2
      5302541.73     15927563.94      5302823.95     15927638.39
#Sta/Elev= 21
       0  40.955  38.632  37.008  70.361  32.546  71.158  31.014  80.617  27.556
  89.957  27.736  96.581  27.356 103.228  27.802 109.829  28.645 116.329  28.747
 128.176  29.731 133.999  32.671 152.884  34.347 172.743  34.426 199.701  34.117
 234.705  35.394 262.306   41.66 274.869  42.844 280.446  45.302 280.643  48.117
 292.192  48.022
#Mann= 3 , 0 , 0
       0    .035       0       0    .035       0 292.192    .035       0
Bank Sta=0,292.192
XS Rating Curve= 0
Exp/Cntr=.3,.1

Type RM Length L Ch R = 1 ,450.2   ,65.617,65.617,65.617
XS GIS Cut Line= 3
      5302523.23      15927637.5      5302675.43     15927679.04
      5302675.43     15927679.04
#Sta/Elev= 17
       0    40.4   6.528  40.728   8.443  44.249  13.896  37.415   38.95  33.537
  50.016  30.721   55.84  29.386  61.654  29.022  69.314  29.442  77.615  29.626
  84.738  29.914  92.402  30.033 106.978  31.607 125.965  34.639  147.06  36.381
  157.92  42.507  157.92  45.801
#Mann= 3 , 0 , 0
       0    .035       0       0    .035       0  157.92    .035       0
Bank Sta=0,157.92
XS Rating Curve= 0
Exp/Cntr=.3,.1

Type RM Length L Ch R = 3 ,450.1   ,,,
BEGIN DESCRIPTION:
A11
END DESCRIPTION:
Bridge Culvert--1,0,-1,-1, 0
Deck Dist Width WeirC Skew NumUp NumDn MinLoCord MaxHiCord MaxSubmerge Is_Ogee
1.64,62.336,2.61,0, 27, 27, , , .95, 0, 0,0,,
       0  38.615  46.752  46.752  50.033  50.033  70.341   71.03  80.446  89.764
  96.391 106.988 106.988 110.269 110.269 116.109 127.953  133.76 152.657 172.507
 199.475 234.449 262.041 274.573 280.151 280.315 291.896
  47.999  47.999  47.999  47.999  47.999  47.999  47.999  47.999  47.999  47.999
  47.999  47.999  47.999  47.999  47.999  47.999  47.999  47.999  47.999  47.999
  47.999  47.999  47.999  47.999  47.999  47.999  47.999
  45.801  45.801  45.801   30.84  30.709  45.801  45.801  45.801  45.801  45.801
  45.801  45.801  31.594  31.824  45.801  45.801  45.801  45.801  45.801  45.801
  45.801  45.801  45.801  45.801  45.801  45.801  45.801
       0  38.615  46.752  46.752  50.033  50.033  70.341   71.03  80.446  89.764
  96.391 106.988 106.988 110.269 110.269 116.109 127.953  133.76 152.657 172.507
 199.475 234.449 262.041 274.573 280.151 280.315 291.896
  47.999  47.999  47.999  47.999  47.999  47.999  47.999  47.999  47.999  47.999
  47.999  47.999  47.999  47.999  47.999  47.999  47.999  47.999  47.999  47.999
  47.999  47.999  47.999  47.999  47.999  47.999  47.999
  45.801  45.801  45.801   30.84  30.709  45.801  45.801  45.801  45.801  45.801
  45.801  45.801  31.594  31.824  45.801  45.801  45.801  45.801  45.801  45.801
  45.801  45.801  45.801  45.801  45.801  45.801  45.801
BR Coef=-1 , 0 , 0 ,1.25, 0 ,,,.8,-1,2,0,
WSPro=,,,, 1 ,,,, 0 ,,,, 0 ,,,,-1 ,-1 ,-1 , 0 , 0 , 0 , 0 , 0
BC Design=,, 0 ,, 0 ,,,,,,
BC HTab Sub Flow Pts= 40
