HEC-RAS study ozz_def.prj: ozzeri

--- ozz_def.g04 (geometry) --- (continued)

Storage Area=c22             ,5319689.3914447,15921717.7674938
Storage Area Surface Line= 6
 5319136.767342315921695.8813908               .
 5319366.571424515921449.6627312               .
 5320138.056557615921613.8085042               .
 5320302.202330715921909.2708957               .
 5320088.812825715921942.1000503               .
 5319103.938187715921695.8813908               .
Storage Area Type= 1
Storage Area Vol Elev= 6
   32.79       0   36.07     .55   39.34   16.33   42.62   54.15    45.9    93.2
   49.18  132.35

Connection=hc_02_04        ,5305765.6462295,15926031.5608869
Connection Line= 4
 5305924.876327915925950.6197587 5305726.805428815926044.8947128
 5305509.816039415926085.9467595 5305525.754123815926079.9697853
Connection Up SA=c04
Connection Dn SA=c02
Conn Weir Coef=3
Conn Weir Is Ogee= 0
Conn Weir SE= 6
       0   49.18      10   49.18      10   43.93     239   43.93     239   49.18
     249   49.18
Connection Culv=1,.1,,10,.035,1,1,1,1,40,40, 1 ,Culvert #1  , 0 ,
     100     100
Conn Culv Bottom n=.035
Conn HTab HWMax=50

Connection=hc_01_03        ,5305617.0666995,15926851.5770318
Connection Line= 4
 5305677.633682815926873.5912814 5305676.473376815926872.8918591
 5305558.552983115926830.7774328 5305555.606755515926829.0475538
Connection Up SA=c03
Connection Dn SA=c01
Conn Weir WD=10
Conn Weir Coef=3
Conn Weir Is Ogee= 0
Conn Weir SE= 6
       0   49.18      10   49.18      10   40.66   501.8   40.66   501.8   49.18
   511.8   49.18
Conn HTab HWMax=50

Connection=hc_03_05        ,5306205.094611,15926812.1797886
Connection Line= 4
 5306232.870135915926798.3418187   5306240.8066915926788.6630064
 5306173.423607815926830.7774328 5306173.278010415926830.9368966
Connection Up SA=c05
Connection Dn SA=c03
Conn Weir WD=10
Conn Weir Coef=3
Conn Weir Is Ogee= 0
Conn Weir SE= 6
       0   49.18      10   49.18      10   39.67  993.61   39.67  993.61   49.18
 1003.61   49.18
Conn HTab HWMax=50

Connection=hc_01_05        ,5305818.9335043,15926549.0864291
Connection Line= 4
   5306011.2810115926520.4470106  5306021.81167315926519.1306777
   5305617.5131815926578.0908746 5305625.128154315926578.6771533
Connection Up SA=c05
Connection Dn SA=c01
Conn Weir WD=10
Conn Weir Coef=3
Conn Weir Is Ogee= 0
Conn Weir SE= 6
       0   49.18      10   49.18      10   43.28   75.57   43.28   75.57   49.18
   85.57   49.18
Conn HTab HWMax=50

Connection=hc_05_07        ,5309325.2871833,15925478.866708
Connection Line= 4
 5309369.182064715925463.9020157 5309380.706467815925460.6092557
 5309279.631844515925494.3007968 5309271.628356415925496.6547639
Connection Up SA=c07
Connection Dn SA=c05
Conn Weir WD=10
Conn Weir Coef=3
Conn Weir Is Ogee= 0
Conn Weir SE= 6
       0   49.18      10   49.18      10   39.67     829   39.67     829   49.18
     839   49.18
Conn HTab HWMax=50

Connection=hc_07_09        ,5313058.990266,15925235.5722775
Connection Line= 4
 5313121.942458315925220.0976842 5313128.890413315925216.3455828
 5312994.124248915925250.0371239 5312991.003943615925255.8087193
Connection Up SA=c09
Connection Dn SA=c07
Conn Weir WD=10
Conn Weir Coef=3
Conn Weir Is Ogee= 0
Conn Weir SE= 6
       0   49.18      10   49.18      10   35.08     665   35.08     665   49.18
     675   49.18
Conn HTab HWMax=50

Connection=hc_09_11        ,5313774.2597862,15924142.1406337
Connection Line= 4
 5313831.077825715924126.5856521 5313836.112329815924125.0534005
 5313709.769050815924158.7449416 5313720.079938615924158.1785408
Connection Up SA=c11
Connection Dn SA=c09
Conn Weir WD=10
Conn Weir Coef=3
Conn Weir Is Ogee= 0
Conn Weir SE= 6
       0   49.18      10   49.18      10   39.34      92   39.34      92   49.18
     102   49.18
Conn HTab HWMax=50

Connection=hc_11_13        ,5315803.2363738,15923205.073318
Connection Line= 4
 5315851.878836815923180.5068101 5315849.181909615923181.6902502
 5315748.107286315923232.2275618 5315763.777462515923225.8686497
Connection Up SA=c13
Connection Dn SA=c11
Conn Weir WD=10
Conn Weir Coef=3
Conn Weir Is Ogee= 0
Conn Weir SE= 6
       0   49.18      10   49.18      10   41.31     993   41.31     993   49.18
    1003   49.18
Conn HTab HWMax=50

Connection=hc_13_15        ,5318221.6707179,15922147.0921544
Connection Line= 4
 5318269.969868515922206.3409408 5318281.6402737 15922218.625686
 5318155.296994615922067.0137512 5318179.775734915922096.3882395
Connection Up SA=c15
Connection Dn SA=c13
Conn Weir WD=10
Conn Weir Coef=3
Conn Weir Is Ogee= 0
Conn Weir SE= 6
       0   49.18      10   49.18      10   34.43     993   34.43     993   49.18
    1003   49.18
Conn HTab HWMax=50

Connection=hc_06_08        ,5309106.0375957,15924848.7771149
Connection Line= 4
 5309183.043855515924823.0614604 5309180.0122542 15924824.152878
 5309028.400319415924874.6901896 5309032.693953615924873.2039316
Connection Up SA=c08
Connection Dn SA=c06
Conn Weir WD=10
Conn Weir Coef=3
Conn Weir Is Ogee= 0
Conn Weir SE= 6
       0   49.18      10   49.18      10   42.62      43   42.62      43   49.18
      53   49.18
Conn HTab HWMax=50

Connection=hc_08_10        ,5311428.1777111,15923737.918387
Connection Line= 4
 5311449.955158315923722.0257432 5311454.191277415923720.7549075
 5311403.653965715923754.4464486 5311404.910443115923754.4464486
Connection Up SA=c10
Connection Dn SA=c08
Conn Weir WD=10
Conn Weir Coef=3
Conn Weir Is Ogee= 0
Conn Weir SE= 6
       0   49.18      10   49.18      10   42.62      43   42.62      43   49.18
      53   49.18
Conn HTab HWMax=50

Connection=hc_10_12        ,5314026.5188721,15922525.8401623
Connection Line= 4
 5314099.483778615922512.1519791 5314105.644658515922513.4266705
 5313945.609838415922538.6953263 5313955.337213115922539.0866732
Connection Up SA=c12
Connection Dn SA=c10
Conn Weir WD=10
Conn Weir Coef=3
Conn Weir Is Ogee= 0
Conn Weir SE= 6
       0   49.18      10   49.18      10   40.98      43   40.98      43   49.18
      53   49.18
Conn HTab HWMax=50

Connection=hc_16_18        ,5315427.1479883,15920683.9294089
Connection Line= 4
 5315406.521840515920634.3544983  5315402.52837315920629.4626547
 5315444.6427993 15920730.537278 5315454.898940315920741.3632046
Connection Up SA=c16
Connection Dn SA=c18
Conn Weir WD=10
Conn Weir Coef=3
Conn Weir Is Ogee= 0
Conn Weir SE= 6
       0   49.18      10   49.18      10   41.97     666   41.97     666   49.18
     676   49.18
Conn HTab HWMax=50

Connection=hc_18_20        ,5315801.6977717,15921643.0274943
Connection Line= 4
 5315747.840450415921572.7885334 5315747.866669115921572.8258051
 5315857.364177615921716.0148547 5315853.719789815921710.4807843
Connection Up SA=c18
Connection Dn SA=c20
Conn Weir WD=10
Conn Weir Coef=3
Conn Weir Is Ogee= 0
Conn Weir SE= 6
       0   49.18      10   49.18      10   41.31     273   41.31     273   49.18
     283   49.18
Conn HTab HWMax=50

Connection=hc_14_20        ,5315342.9698449,15922083.6579809
Connection Line= 4
 5315287.910655315922108.6979363 5315275.246726715922114.5608581
 5315414.365758115922051.1389467 5315394.356239515922060.2341825
Connection Up SA=c14
Connection Dn SA=c20
Conn Weir WD=10
Conn Weir Coef=3
Conn Weir Is Ogee= 0
Conn Weir SE= 6
       0   49.18      10   49.18      10   33.77      76   33.77      76   49.18
      86   49.18
Conn HTab HWMax=50

Connection=hc_14_18        ,5315169.1134249,15921698.5175615
Connection Line= 4
 5315113.396569715921731.7474552 5315095.210333115921740.1669942
 5315254.788045615921650.1487974 5315213.058751315921672.0069992
Connection Up SA=c14
Connection Dn SA=c18
Conn Weir WD=10
Conn Weir Coef=3
Conn Weir Is Ogee= 0
Conn Weir SE= 6
       0   49.18      10   49.18      10   36.07     174   36.07     174   49.18
     184   49.18
Conn HTab HWMax=50

Connection=hc_14_16        ,5314805.435288,15920887.3562974
Connection Line= 4
 5314743.216720815920932.1589966 5314724.9082054 15920940.635164
 5314892.669390315920830.1582861 5314860.946835615920846.4727429
Connection Up SA=c14
Connection Dn SA=c16
Conn Weir WD=10
Conn Weir Coef=3
Conn Weir Is Ogee= 0
Conn Weir SE= 6
       0   49.18      10   49.18      10   36.07     174   36.07     174   49.18
     184   49.18
Conn HTab HWMax=50

Chan Stop Cuts=-1

--- ozz_def.g01 (geometry) ---

Geom Title=studio_ozz
Version=Version 3.0.1  Mar 2001

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
River Reach=OZZERI          ,tronco_1

--- ozz_def.g02 (geometry) ---

Geom Title=studio_ozz_mod
Version=Version 3.0.1  Mar 2001

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
River Reach=OZZERI          ,tronco_1
Reach XY= 30
      1621737.73      4853081.72      1621077.53      4852982.57
      1620854.84      4852876.29      1620679.28      4852906.77
      1620557.84      4853099.24      1620266.19      4853092.11
      1620045.62       4853207.6       1619658.9      4853315.14
      1619452.34      4853558.01      1619256.33        4853606.
      1619083.93      4853536.01       1618903.9      4853650.49
      1618714.74       4853688.6      1618397.51      4853993.23
      1617877.88      4854119.85      1617682.12      4854377.78
      1617497.89      4854423.77      1617225.88      4854345.75
      1616607.94      4854537.07      1616227.23      4854748.73
      1616196.06      4854844.88      1616064.04      4854962.02
      1615357.05      4854693.79      1614782.97      4854356.77
      1614219.36      4853925.94       1613501.3       4851973.5
      1612807.86      4850902.43      1613320.95      4850272.55
      1613997.96      4849717.94      1614042.97      4849561.47

Type RM Length L Ch R = 1 ,850     ,58.8,58.8,58.8
XS GIS Cut Line= 4
      1621711.17      4853038.08        1621685.      4853074.38
  1621684.999942 4853074.3800805 1621684.9981893 4853074.3825132
#Sta/Elev= 16
       0  11.798   9.915  11.798  13.277  11.695  15.081  11.057   17.59  10.816
  18.218   10.06  19.874   9.986  21.811   9.665   23.77    9.59   25.34   9.893
  26.005  10.415  28.342   11.31  30.323  12.045  34.268  12.174  36.085  11.911
  44.773   11.76
#Mann= 3 , 0 , 0
       0    .035       0       0    .035       0  44.773    .035       0
Bank Sta=0,44.773
XS Rating Curve= 0
Exp/Cntr=.3,.1

Type RM Length L Ch R = 1 ,849     ,75.65,75.65,75.65
XS GIS Cut Line= 2
       1621639.9      4853014.01  1621642.329941  4853059.188903
#Sta/Elev= 14
       0  12.095   9.884  12.181  17.617  12.143  21.578  10.575  22.088  10.112
  23.868   9.955  26.057   9.717  28.155   9.801  29.998   9.995  30.865  10.731
  34.856  12.183  37.986  12.492  41.366  12.351  45.379  12.004
#Mann= 3 , 0 , 0
       0    .035       0       0    .035       0  45.379    .035       0
Bank Sta=0,45.379
XS Rating Curve= 0
Exp/Cntr=.3,.1

Type RM Length L Ch R = 1 ,848     ,26.45,26.45,26.45
XS GIS Cut Line= 2
      1621567.25      4853037.89 1621570.4896093 4853071.7359179
#Sta/Elev= 17
       0  10.733   2.913  10.702   3.163  11.854  11.314  12.084  12.448   10.63
  15.516  10.523  16.282  10.121  17.789   9.969  19.748   9.505  21.675   9.693
    22.8   9.801  23.941   9.919  24.712  10.579  26.628  11.177   28.98  12.051
  32.292  12.404  34.256  12.284
#Mann= 3 , 0 , 0
       0    .035       0       0    .035       0  34.256    .035       0
Bank Sta=0,34.256
XS Rating Curve= 0
Exp/Cntr=.3,.1

Type RM Length L Ch R = 1 ,847     ,41.47,41.47,41.47
XS GIS Cut Line= 3
      1621541.88       4853037.1      1621541.11      4853077.97
 1621541.1099454 4853077.9728987
#Sta/Elev= 17
       0  11.886   9.401  12.065   14.06  12.102   16.57  11.071  19.151   10.59
  19.877  10.077  21.336    9.82  23.278   9.496  25.528   9.624  27.142   9.929
   28.43  10.234  31.281  10.209  31.645   11.69  33.594  11.911  35.689  11.973
  35.777  10.196  40.943   10.15
#Mann= 3 , 0 , 0
       0    .035       0       0    .035       0  40.943    .035       0
Bank Sta=0,40.943
XS Rating Curve= 0
Exp/Cntr=.3,.1

Type RM Length L Ch R = 1 ,846     ,97.85,97.85,97.85
XS GIS Cut Line= 2
      1621502.64      4853038.49 1621499.2905587  4853067.675132
#Sta/Elev= 14
       0  10.714   5.276  10.674   5.563   11.88   8.591  11.659   9.556  10.921
  13.107  10.169  15.284   9.886  16.718   9.584  18.842   9.523  20.354   9.645
  21.211  10.361   23.59  11.153  25.611  11.992  29.415  12.069
#Mann= 3 , 0 , 0
       0    .035       0       0    .035       0  29.415    .035       0
Bank Sta=0,29.415
XS Rating Curve= 0
Exp/Cntr=.3,.1

Type RM Length L Ch R = 1 ,845     ,61.95,61.95,61.95
XS GIS Cut Line= 2
      1621404.92      4853027.46 1621403.6702072  4853058.194904
#Sta/Elev= 17
       0  11.824   3.296  11.644   4.257  11.072    6.09  10.703   6.824   10.04
   8.756   9.606  10.826   9.606  12.869   9.813  14.466   9.815  15.139   9.895
  15.296  10.289  18.707  10.192  18.827  11.398  19.507  11.709   23.08  11.886
  23.193  10.182  30.865  10.323
#Mann= 3 , 0 , 0
       0    .035       0       0    .035       0  30.865    .035       0
Bank Sta=0,30.865
XS Rating Curve= 0
Exp/Cntr=.3,.1

Type RM Length L Ch R = 1 ,844     ,64.8,64.8,64.8
XS GIS Cut Line= 2
      1621348.22      4853001.51 1621339.9703435 4853046.3881316
#Sta/Elev= 17
       0  11.597  12.908  11.688  15.127  11.527  16.103  12.115  18.006  12.239
  20.212   11.32  22.696  10.528   23.11    9.96  25.131   9.832  27.281   9.714
  29.755   9.874  31.566   9.855  33.165    11.1  35.805  12.196  37.637  12.138
  39.545  11.909  45.708  11.635
#Mann= 3 , 0 , 0
       0    .035       0       0    .035       0  45.708    .035       0
Bank Sta=0,45.708
XS Rating Curve= 0
Exp/Cntr=.3,.1

Type RM Length L Ch R = 1 ,843     ,56.1,56.1,56.1
XS GIS Cut Line= 2
      1621284.39      4852998.35 1621275.1904244 4853038.4881483
#Sta/Elev= 16
       0  10.792   7.467  10.708   7.658  12.149  10.218  12.048   11.91  11.403
  12.322  10.683  15.345  10.098  17.414   9.853   19.33    9.65   21.84   9.837
   23.87  10.002  25.421  11.047  28.406   12.13  31.384  12.282  33.581  11.796
  41.268  11.583
#Mann= 3 , 0 , 0
       0    .035       0       0    .035       0  41.268    .035       0
Bank Sta=0,41.268
XS Rating Curve= 0
Exp/Cntr=.3,.1

Type RM Length L Ch R = 1 ,842     ,64.59,64.59,64.59
XS GIS Cut Line= 2
      1621227.82      4852983.93      1621220.32      4853031.92
#Sta/Elev= 15
       0  11.985   9.606  11.932  16.281  11.568  18.542  10.808  19.409   9.957
   21.16   9.676  23.349   9.657  26.015  10.039  27.215  10.117  28.685   10.11
  29.736  10.716  32.932  12.204  36.046  12.125  38.107  11.599   48.59  11.611
#Mann= 3 , 0 , 0
       0    .035       0       0    .035       0   48.59    .035       0
Bank Sta=0,48.59
XS Rating Curve= 0
Exp/Cntr=.3,.1

Type RM Length L Ch R = 1 ,841     ,83.78,83.78,83.78
XS GIS Cut Line= 2
      1621160.89      4852974.87 1621160.7600139  4853020.705102
#Sta/Elev= 14
       0  12.296  13.362  12.199  15.445  11.164  16.675  10.126  19.206   9.477
  21.261   9.106  23.813   9.979  24.962   9.672  28.225  10.143  32.616  10.362
  32.659  12.777   34.27  12.824  34.454  10.217  45.965  10.314
#Mann= 3 , 0 , 0
       0    .035       0       0    .035       0  45.965    .035       0
Bank Sta=0,45.965
XS Rating Curve= 0
Exp/Cntr=.3,.1

Type RM Length L Ch R = 1 ,840     ,60.15,60.15,60.15
XS GIS Cut Line= 2
      1621086.76      4852954.73 1621065.3800346  4853014.659903
#Sta/Elev= 17
       0  13.868  10.525  13.809  14.172  11.699  20.225  10.686  21.053  10.028
  22.298   9.777  26.205    9.75  29.343   9.706  31.819   9.875  33.532  10.076
  34.585  10.256  35.652  10.763  38.229  11.056  41.817  13.075  44.615  13.026
  47.518   12.18   63.69  12.138
#Mann= 3 , 0 , 0
       0    .035       0       0    .035       0   63.69    .035       0
Bank Sta=0,63.69
XS Rating Curve= 0
Exp/Cntr=.3,.1

Type RM Length L Ch R = 1 ,839     ,65.63,65.63,65.63
XS GIS Cut Line= 3
       1621042.3      4852920.91      1621009.79      4852983.32
 1621009.7886113  4852983.322666
#Sta/Elev= 20
       0  13.469  10.298  13.602  11.295  13.051  11.976  12.951  12.941  13.592
  23.454  13.067  26.308  11.223  30.145  10.642  33.173   10.05  34.705   9.812
  36.881   9.773  39.113   9.887  42.591  10.065   46.14  10.255  46.711  10.513
  49.976  10.981  53.596  12.986  58.662  12.986  62.418   12.53  70.563  12.586
#Mann= 3 , 0 , 0
       0    .035       0       0    .035       0  70.563    .035       0
Bank Sta=0,70.563
XS Rating Curve= 0
Exp/Cntr=.3,.1

Type RM Length L Ch R = 1 ,838.5   ,9.4,9.4,9.4
XS GIS Cut Line= 3
      1620983.82      4852891.82      1620961.33      4852935.82
 1620961.3294982 4852935.8209817
#Sta/Elev= 19
       0  13.371   6.516   13.49  15.508  13.544  17.391  13.057  19.705  11.711
  20.856   10.74  23.588  10.704  24.247  10.462  25.204  10.074  27.838   9.406
  30.964   9.263  32.517   9.342  33.584   9.397  38.188   9.812  38.766  10.072
  39.787  10.453  43.211  11.036  46.631  11.161  49.671    9.83
#Mann= 3 , 0 , 0
       0    .035       0       0    .035       0  49.671    .035       0
Bank Sta=0,49.671
XS Rating Curve= 0
Exp/Cntr=.3,.1

Type RM Length L Ch R = 1 ,838     ,18.51,18.51,18.51
XS GIS Cut Line= 2
      1620975.23      4852890.33 1620946.3383299 4852936.7050883
#Sta/Elev= 19
       0  13.364  12.542  13.645  19.061  13.908  19.515  10.811   21.65  10.545
  21.983  10.152  24.848   9.781  26.617   9.579  28.686   9.744  30.654   9.682
  33.005   9.884  36.211  10.101  38.517  10.798  38.523  14.033  44.664  14.006
  44.702  13.378  46.563  13.392  49.993  12.088  55.587  11.993
#Mann= 3 , 0 , 0
       0    .035       0       0    .035       0  55.587    .035       0
Bank Sta=0,55.587
XS Rating Curve= 0
Exp/Cntr=.3,.1

Type RM Length L Ch R = 1 ,837.5   ,34.4,34.4,34.4
XS GIS Cut Line= 3
      1620959.81       4852879.7      1620928.26      4852929.13
 1620928.2599466 4852929.1300836
#Sta/Elev= 25
       0  13.248    6.83  13.488  10.048  13.434  10.989  13.749  12.023  13.848
  13.729  13.514  17.894  11.093   21.57  10.598  22.076  10.097  23.319    9.63
  23.912   9.595   25.76   9.203  27.877   9.095  30.335   9.128  32.086   9.289
  34.371   9.593  35.014   9.826  35.186  10.095  36.535  10.407  39.685  10.823
  43.751  12.932  44.855   13.22  48.912  13.286  51.226  12.752    58.8  12.099
#Mann= 3 , 0 , 0
       0    .035       0       0    .035       0    58.8    .035       0
Bank Sta=0,58.8
XS Rating Curve= 0
Exp/Cntr=.3,.1

Type RM Length L Ch R = 1 ,837     ,61.54,61.54,61.54
XS GIS Cut Line= 3
      1620927.75       4852861.5      1620900.54       4852916.2
 1620900.5395549 4852916.2008949
#Sta/Elev= 19
       0  12.858   9.689   12.91  14.378  12.782  15.688  12.483   18.47  10.989
   21.99  10.545  22.651   10.28  22.852  10.133  25.683   9.682  28.265   9.565
  30.174   9.623  31.516   9.727    34.6   10.19  35.603  10.583  39.488  11.091
   42.46  13.018   47.79  13.151  50.373  12.297  61.111  12.122
#Mann= 3 , 0 , 0
       0    .035       0       0    .035       0  61.111    .035       0
Bank Sta=0,61.111
XS Rating Curve= 0
Exp/Cntr=.3,.1

Type RM Length L Ch R = 1 ,798     ,52.98,52.98,52.98
XS GIS Cut Line= 3
      1620853.37      4852847.09       1620856.3       4852905.3
 1620856.3001962 4852905.3038975
#Sta/Elev= 19
       0  13.852    8.97  13.858   13.23  13.767  16.492   12.29  17.386  11.351
  23.585  10.848  24.414  10.466  24.581  10.043  26.846   9.668  29.263   9.568
  31.228   9.713  33.433   9.816  35.519   10.15  36.641  10.704  40.488  10.955
  44.261  12.762  48.207  12.777  50.311   12.32  58.324  12.379
#Mann= 3 , 0 , 0
       0    .035       0       0    .035       0  58.324    .035       0
Bank Sta=0,58.324
XS Rating Curve= 0
Exp/Cntr=.3,.1

Type RM Length L Ch R = 1 ,797     ,87.49,87.49,87.49
XS GIS Cut Line= 3
      1620801.07      4852848.01      1620803.37      4852913.55
 1620803.3701086 4852913.5530956
#Sta/Elev= 22
       0  13.329  12.412  13.603  16.847  13.542  20.836  11.431   26.26  10.917
  27.345  10.501  27.622  10.143  30.702   9.592  32.834   9.394  34.818   9.746
  36.734   9.945  38.469   9.868  40.104  11.017  43.531  11.078  47.312  13.152
  50.461  13.161  52.198  12.783  53.887   12.92  55.019  13.239  57.016  13.138
  58.656  12.557  65.643  12.062
#Mann= 3 , 0 , 0
       0    .035       0       0    .035       0  65.643    .035       0
Bank Sta=0,65.643
XS Rating Curve= 0
Exp/Cntr=.3,.1

Type RM Length L Ch R = 1 ,796     ,38.51,38.51,38.51
XS GIS Cut Line= 2
      1620711.67      4852871.07 1620719.5993446 4852920.0459519
#Sta/Elev= 17
       0  10.064     .29    11.1   6.721  10.925   9.733   10.83  14.342   10.24
  21.301  10.077  24.219   9.881  25.776   9.679  27.059   9.618  28.663   9.775
  30.617  10.161  32.277  10.742  36.014  10.982  39.545   13.04  42.051  13.377
  45.103  12.632  49.856  12.682
#Mann= 3 , 0 , 0
       0    .035       0     .29    .035       0  49.856    .035       0
Bank Sta=.29,49.856
XS Rating Curve= 0
Exp/Cntr=.3,.1

Type RM Length L Ch R = 1 ,795     ,55.31,55.31,55.31
XS GIS Cut Line= 2
      1620673.78       4852883.3 1620683.2499773 4852923.5999035
#Sta/Elev= 16
       0  13.653   6.262  13.564   9.472  11.602  14.692  10.853  15.616  10.365
  15.989  10.011  17.972   9.921  19.855   9.891  22.075   9.858  24.137   9.681
  27.171  10.079  28.089  10.605  31.799  10.845  36.566  13.136  38.999  13.515
   41.45  12.906
#Mann= 3 , 0 , 0
       0    .035       0       0    .035       0   41.45    .035       0
Bank Sta=0,41.45
XS Rating Curve= 0
Exp/Cntr=.3,.1

Type RM Length L Ch R = 1 ,794     ,98.95,98.95,98.95
XS GIS Cut Line= 2
      1620606.27      4852920.35 1620653.3347179 4852943.7973685
#Sta/Elev= 15
       0  12.772  12.714  12.335  17.097  10.585  21.711  10.086  22.119   9.958
  23.986    9.68  26.368   9.736  29.063    9.87  31.145   9.893  32.959   9.934
  33.998  10.335   39.37  10.888  44.177  13.729   48.19  13.876  52.694  13.298
#Mann= 3 , 0 , 0
       0    .035       0       0    .035       0  52.694    .035       0
Bank Sta=0,52.694
XS Rating Curve= 0
Exp/Cntr=.3,.1

Type RM Length L Ch R = 1 ,793     ,49.41,49.41,49.41
XS GIS Cut Line= 3
       1620587.7       4853028.6      1620635.68      4853032.41
 1620635.6830878 4853032.4102452
#Sta/Elev= 15
       0  12.616   6.719  12.992   8.123  13.457  10.513   13.39  14.112  10.751
  17.036  10.577  17.962   9.975  22.341   9.649  24.345   9.514  29.029   8.892
  32.079  10.262  32.233  10.941  35.396  12.953  45.552  13.032  48.883  13.056
#Mann= 3 , 0 , 0
       0    .035       0   8.123    .035       0  48.883    .035       0
Bank Sta=8.123,48.883
XS Rating Curve= 0
Exp/Cntr=.3,.1

Type RM Length L Ch R = 1 ,792     ,40.36,40.36,40.36
XS GIS Cut Line= 3
      1620567.35      4853049.18      1620606.05      4853091.55
 1620606.0514175  4853091.551552
#Sta/Elev= 19
       0  12.366  12.949  12.593  15.591   13.27  17.787  13.204  21.789  11.296
  25.636    10.8  27.162  10.128  27.378   9.924   29.15   9.658  31.367   9.786
  33.813   9.584  36.046   9.599  39.151   9.547  40.441  10.705  42.756  10.926
  47.592  13.424  50.457  13.649  52.972  12.745  57.442  12.589
#Mann= 3 , 0 , 0
       0    .035       0  15.591    .035       0  50.457    .035       0
Bank Sta=15.591,50.457
XS Rating Curve= 0
Exp/Cntr=.3,.1

Type RM Length L Ch R = 1 ,791     ,45.53,45.53,45.53
XS GIS Cut Line= 2
      1620546.74      4853070.52 1620570.9199644 4853133.2999075
#Sta/Elev= 20
       0  12.418   6.884   12.55   8.455  12.887  12.407  13.009  16.475  11.099
  20.953  10.493   21.86   9.896  23.693   9.725  26.221   9.721  28.086   9.186
   30.82   9.178  33.044   9.836  35.295  10.907  38.584  11.344  42.355  13.563
  45.586  13.502  52.105  13.172   62.96  12.643  64.124  12.077   67.39  11.934
#Mann= 3 , 0 , 0
       0    .035       0  12.407    .035       0  42.355    .035       0
Bank Sta=12.407,42.355
XS Rating Curve= 0
Exp/Cntr=.3,.1

Type RM Length L Ch R = 1 ,790     ,112.03,112.03,112.03
XS GIS Cut Line= 3
      1620509.06      4853082.96      1620518.61      4853146.84
 1620518.6102956 4853146.8419769
#Sta/Elev= 23
       0  12.155   6.127  12.429   7.134  12.678   9.973  12.425  11.868  11.446
  16.758  10.617   18.16   9.931  19.787   9.873  21.747   9.632  23.737   9.457
  26.716   9.289  28.378   9.675  29.466   9.693  30.963  10.631  34.512  10.903
  37.886  13.042  44.889  13.152  47.417  12.109  50.607  11.749  51.171  11.207
   51.72  11.257   52.68  11.777  64.672  11.961
#Mann= 3 , 0 , 0
       0    .035       0   7.134    .035       0  44.889    .035       0
Bank Sta=7.134,44.889
XS Rating Curve= 0
Exp/Cntr=.3,.1

Type RM Length L Ch R = 1 ,788     ,99.84,99.84,99.84
XS GIS Cut Line= 2
      1620410.07      4853081.95 1620393.5507692 4853146.3869995
#Sta/Elev= 21
       0  12.015   9.355  12.538  14.959  12.427  17.753  10.911  21.531  10.564
  22.984  10.019  23.199   9.573   25.47   9.289  27.636    9.44    29.7   9.344
  31.704   9.297  33.881   9.132  35.165   9.707  36.281  10.427   39.79  10.528
  42.894  12.995  47.613  12.721  50.435  10.417  52.704  10.274  53.564  11.408
  66.817  11.551
#Mann= 3 , 0 , 0
       0    .035       0   9.355    .035       0  66.817    .035       0
Bank Sta=9.355,66.817
XS Rating Curve= 0
Exp/Cntr=.3,.1

Type RM Length L Ch R = 1 ,786     ,41.02,41.02,41.02
XS GIS Cut Line= 3
       1620302.9      4853054.54      1620301.53       4853130.7
 1620301.5299838 4853130.7009001
#Sta/Elev= 18
       0  10.423   7.603  10.491   7.881  12.376  10.303  12.605  10.407  10.527
  17.705   9.943  20.695   9.554  22.763   9.536  25.076    9.28  27.016   9.195
  29.024   9.127  31.054   9.026  33.933   9.354  35.575  10.504  39.057  10.819
  42.331  12.684  49.253  12.487  76.741  12.039
#Mann= 3 , 0 , 0
       0    .035       0       0    .035       0  76.741    .035       0
Bank Sta=0,76.741
XS Rating Curve= 0
Exp/Cntr=.3,.1

Type RM Length L Ch R = 1 ,785     ,45.12,45.12,45.12
XS GIS Cut Line= 2
      1620252.58      4853060.95 1620286.8459907 4853140.1907284
#Sta/Elev= 20
       0  12.678  10.981  12.661  16.373  12.871  17.308  12.296  18.072  11.052
  21.961   10.81  22.586  10.499  22.727   9.842   24.89   9.527  27.112    9.51
  29.142   9.466  31.043   9.371   34.07   9.271  35.544   9.571  36.492   9.559
  38.721  11.017   42.29  11.335  44.695   12.94   52.38  12.577   86.44  12.035
#Mann= 3 , 0 , 0
       0    .035       0       0    .035       0   86.44    .035       0
Bank Sta=0,86.44
XS Rating Curve= 0
Exp/Cntr=.3,.1

Type RM Length L Ch R = 1 ,784     ,29.61,29.61,29.61
XS GIS Cut Line= 3
      1620211.99      4853079.74      1620253.08      4853159.96
 1620253.0800487 4853159.9600951
#Sta/Elev= 16
       0  10.728  17.533  10.817  21.454  10.297  26.337  10.245   27.88   9.806
  30.437   9.508  32.967   9.457  34.947    9.46  36.956   9.245  40.482   9.559
  42.682   9.543  44.895  10.991  47.605  11.114  51.452  13.251  56.151  13.058
   90.48   12.19
#Mann= 3 , 0 , 0
       0    .035       0       0    .035       0   90.48    .035       0
Bank Sta=0,90.48
XS Rating Curve= 0
Exp/Cntr=.3,.1

Type RM Length L Ch R = 1 ,783     ,48.88,48.88,48.88
XS GIS Cut Line= 3
      1620180.51      4853096.17      1620214.37      4853147.23
 1620214.3716571 4853147.2324988
#Sta/Elev= 23
       0  13.268  18.082  13.498   18.97  13.685  21.474  13.471  24.341  11.626
  28.484  11.174  29.531  10.545  29.925   9.823   32.21   9.696  35.347   9.401
  38.822   9.325  43.599   9.362  45.334   9.591  54.608   9.481  54.802  13.739
  55.462  13.729  55.496  13.073  57.405  12.983  57.593   9.821  60.301   9.987
  60.416  12.164  61.451  12.145  61.543    9.95
#Mann= 3 , 0 , 0
       0    .035       0       0    .035       0  61.543    .035       0
Bank Sta=0,61.543
XS Rating Curve= 0
Exp/Cntr=.3,.1

Type RM Length L Ch R = 1 ,782     ,37.5,37.5,37.5
XS GIS Cut Line= 3
      1620150.36      4853135.54      1620186.54      4853199.92
 1620186.5410279 4853199.9218291
#Sta/Elev= 19
       0   13.55     .73  13.692    .756  14.197   4.674  13.832   8.136  11.652
  12.101  11.079  13.622   9.704  15.416    9.47   18.93   9.417  20.158   9.409
  22.251   9.455  24.395    9.36   27.42   9.318   29.56   9.628  31.534  10.879
  34.671  10.936  38.717  13.521  43.967  13.544  73.992  12.711
#Mann= 3 , 0 , 0
       0    .035       0     .73    .035       0  43.967    .035       0
Bank Sta=.73,43.967
XS Rating Curve= 0
Exp/Cntr=.3,.1

Type RM Length L Ch R = 1 ,781     ,23.62,23.62,23.62
XS GIS Cut Line= 2
      1620120.18      4853151.24 1620140.4187484 4853195.2972754
#Sta/Elev= 15
       0  14.069   3.286  13.776   6.708  11.595  10.604  11.085  12.015   9.797
  14.412   9.458      17   9.492  20.057   9.205   23.04   9.306  25.222   9.159
  26.635   9.264  28.437   9.514  33.628   9.988  43.604  10.461  49.417  10.656
#Mann= 3 , 0 , 0
       0    .035       0       0    .035       0  49.417    .035       0
Bank Sta=0,49.417
XS Rating Curve= 0
Exp/Cntr=.3,.1

Type RM Length L Ch R = 1 ,780     ,9,9,9
XS GIS Cut Line= 2
      1620098.28      4853160.07 1620110.2993129 4853192.9081229
#Sta/Elev= 16
       0  13.689   2.377  13.597   6.252  11.084    8.97  10.778  10.878   9.765
  12.813   9.876  14.798   9.874  16.574   9.873   19.15   9.876  21.876   9.878
   25.14   9.885  26.838   9.891  28.122   9.513  28.702  10.528  32.225  11.604
  35.228   13.15
#Mann= 3 , 0 , 0
       0    .035       0       0    .035       0  35.228    .035       0
Bank Sta=0,35.228
XS Rating Curve= 0
Exp/Cntr=.3,.1

Type RM Length L Ch R = 3 ,779.5   ,,,
BEGIN DESCRIPTION:
Ponte di Pontetetto
END DESCRIPTION:
Bridge Culvert--1,0,-1,-1, 0
Deck Dist Width WeirC Skew NumUp NumDn MinLoCord MaxHiCord MaxSubmerge Is_Ogee
.5,8,1.44,0, 19, 19, , , .95, 0, 0,0,,
       0    2.37    6.24     7.6    8.96   10.87   12.22   12.85   15.74   16.56
   19.13   21.85   22.28    25.1   26.59   27.88   28.45   32.23   35.23
      14      14      14      14      14      14      14      14      14      14
      14      14      14      14      14      14      14      14      14
   13.69    13.6   11.08   12.75   13.08   12.69   12.31    9.52    9.37    12.3
   12.96   11.69    9.37     9.3   12.48   12.93      13    11.6   13.15
       0    2.37    6.24     7.6    8.96   10.87   12.22   12.85   15.74   16.56
   19.13   21.85   22.28    25.1   26.59   27.88   28.45   32.23   35.23
      14      14      14      14      14      14      14      14      14      14
      14      14      14      14      14      14      14      14      14
   13.69    13.6   11.08   12.75   13.08   12.69   12.31    9.52    9.37    12.3
   12.96   11.69    9.37     9.3   12.48   12.93      13    11.6   13.15
BR Coef=-1 , 0 , 0 ,1.25, 0 ,,,.8,-1,2,0,
WSPro=,,,, 1 ,,,, 0 ,,,, 0 ,,,,-1 ,-1 ,-1 , 0 , 0 , 0 , 0 , 0
BC Design=,, 0 ,, 0 ,,,,,,
BC HTab Sub Flow Pts= 40

Type RM Length L Ch R = 1 ,779.3   ,9.1,9.1,9.1
XS GIS Cut Line= 2
      1620098.28      4853160.07 1620110.2993129 4853192.9081229
#Sta/Elev= 16
       0  13.689   2.377  13.597   6.252  11.084    8.97  10.778  10.878   9.765
  12.813   9.876  14.798   9.874  16.574   9.873   19.15   9.876  21.876   9.878
   25.14   9.885  26.838   9.891  28.122   9.513  28.702  10.528  32.225  11.604
  35.228   13.15
#Mann= 3 , 0 , 0
       0    .035       0       0    .035       0  35.228    .035       0
Bank Sta=0,35.228
XS Rating Curve= 0
Exp/Cntr=.3,.1

Type RM Length L Ch R = 1 ,779     ,19.07,19.07,19.07
XS GIS Cut Line= 3
      1620088.08      4853157.61      1620102.44      4853197.85
 1620102.4406398 4853197.8517928
#Sta/Elev= 14
       0  11.508   5.706  13.242   5.736  14.151   6.132  14.156    6.37   9.994
  11.452  10.093  20.922   9.658  23.684   9.273  27.048   9.566  31.138   9.462
   32.88   9.569  34.034  10.557  39.263  11.387  42.872  13.546
#Mann= 3 , 0 , 0
       0    .035       0       0    .035       0  42.872    .035       0
Bank Sta=0,42.872
XS Rating Curve= 0
Exp/Cntr=.3,.1

Type RM Length L Ch R = 1 ,778.5   ,37.61,37.61,37.61
XS GIS Cut Line= 2
      1620072.65      4853168.62 1620083.6699726 4853206.8999047
#Sta/Elev= 21
       0  14.249     .07  13.162   4.641  13.075   6.297  11.547  10.179  11.299
   11.84  10.476  12.647   9.815    14.2   9.106  17.562   8.961  22.099   8.995
  24.974   8.904  27.337   9.392  27.885   9.805  30.525  11.225  33.551  11.282
  36.587  13.139  37.548  13.376  39.522  13.614  39.633  13.851   39.87  13.862
   39.99  12.967
#Mann= 3 , 0 , 0
       0    .035       0       0    .035       0   39.99    .035       0
Bank Sta=0,39.99
XS Rating Curve= 0
Exp/Cntr=.3,.1

Type RM Length L Ch R = 1 ,778     ,45.47,45.47,45.47
XS GIS Cut Line= 2
      1620034.46      4853174.11  1620065.606733 4853265.1604497
#Sta/Elev= 19
       0  13.335   8.221  13.344  11.964  13.282  14.126  11.527  17.365  11.406
   19.28  10.503  19.737   9.716  21.866   9.684  24.775   9.539  27.244    9.64
  30.218   9.539  33.361   9.445  35.356   9.383   36.32  10.354  39.461  11.802
  44.566  13.433  47.004  13.613  49.438  13.037    96.3  12.739
#Mann= 3 , 0 , 0
       0    .035       0       0    .035       0    96.3    .035       0
Bank Sta=0,96.3
XS Rating Curve= 0
Exp/Cntr=.3,.1

Type RM Length L Ch R = 1 ,777     ,52.65,52.65,52.65
XS GIS Cut Line= 2
      1619991.09      4853183.58  1620016.289971 4853266.0099052
#Sta/Elev= 18
       0  13.418  16.654  13.332  19.299   11.62  23.238  11.313  25.494   9.844
  27.163   9.437  30.173   9.733  32.417    9.64  36.384   9.631  38.746   9.421
  40.978   9.315  41.747  10.025   44.61  11.764  47.475  11.932  49.818  13.315
  52.293  13.585  53.267  12.923    86.4  12.601
#Mann= 3 , 0 , 0
       0    .035       0       0    .035       0    86.4    .035       0
Bank Sta=0,86.4
XS Rating Curve= 0
Exp/Cntr=.3,.1

Type RM Length L Ch R = 1 ,776     ,106.06,106.06,106.06
XS GIS Cut Line= 2
      1619940.14      4853207.27  1619946.380491  4853222.750555
#Sta/Elev= 18
       0  13.687   4.782  13.878  10.701  13.792  13.697  11.876  17.643  11.513
  20.323   9.844  22.918   9.695   25.04   9.695  29.016   9.697  33.095   9.527
  35.555   9.405  36.222  10.133  39.203  11.579  42.657  11.863  45.136  13.197
  46.788  13.382  48.438  12.359   80.16   12.42
#Mann= 3 , 0 , 0
       0    .035       0       0    .035       0   80.16    .035       0
Bank Sta=0,80.16
XS Rating Curve= 0
Exp/Cntr=.3,.1

Type RM Length L Ch R = 1 ,775     ,3.39,3.39,3.39
XS GIS Cut Line= 3
      1619840.75      4853245.42      1619915.65      4853267.55
 1619915.6510536 4853267.5503113
#Sta/Elev= 20
       0  13.777   5.114  13.693   6.399  13.444   9.337  13.328  11.797  11.823
  15.749   11.42  18.534   9.877  18.725   9.592  21.054   9.382  25.291   9.342
  28.708   9.212  31.866   9.223  33.932   9.167  35.039  10.047  38.357  11.659
  40.913  11.732  43.694  13.054  45.378  13.098  47.526  12.471  56.291  12.391
#Mann= 3 , 0 , 0
       0    .035       0       0    .035       0  43.694    .035       0
Bank Sta=0,43.694
XS Rating Curve= 0
Exp/Cntr=.3,.1

Type RM Length L Ch R = 1 ,774     ,70.95,70.95,70.95
XS GIS Cut Line= 2
      1619843.51      4853219.32      1619854.09      4853311.96
#Sta/Elev= 19
       0  14.053   7.625  13.727  17.579  10.707  29.361  10.305  31.605   9.876
  40.062   9.649  44.514    9.72  48.179   9.402  51.367   9.405  53.772   9.309
  55.499    9.24  57.188   9.651  60.044  11.498   63.61  11.786   66.73  13.447
  69.989  13.602   73.06  13.076   83.59  12.635   93.37  12.161
#Mann= 3 , 0 , 0
       0    .035       0       0    .035       0   93.37    .035       0
Bank Sta=0,93.37
XS Rating Curve= 0
Exp/Cntr=.3,.1

Type RM Length L Ch R = 1 ,773     ,68.49,68.49,68.49
XS GIS Cut Line= 3
      1619772.16      4853246.71      1619789.45      4853325.24
 1619789.4508613 4853325.2439117
#Sta/Elev= 18
       0  13.272  18.176  13.404  20.055  12.978  23.472  11.443  27.592  10.875
   29.44  10.068  29.661   9.744   32.11   9.611  35.157   9.547  38.472   9.552
  42.046    9.31  45.288   9.449  47.846   9.588  49.181  10.963  52.615  11.332
  55.672  13.155  64.143  12.999  80.424  12.879
#Mann= 3 , 0 , 0
       0    .035       0       0    .035       0  80.424    .035       0
Bank Sta=0,80.424
XS Rating Curve= 0
Exp/Cntr=.3,.1

Type RM Length L Ch R = 1 ,772.5   ,12.3,12.3,12.3
#Sta/Elev= 27
       0  16.206   6.349  16.704  11.854  16.606  14.312  14.821  16.425  13.136
    18.1  12.998  20.904  11.312  24.939  11.132  27.027  10.125  27.608   9.769
  28.206    9.46  29.948   9.396  30.942   8.855  33.627   8.495  36.539   8.397
  39.521   8.375  42.037   8.312   44.24    9.35  44.693   9.531  45.042   9.765
  46.736  11.054   46.77  11.042  50.482  11.671  53.461  13.415   55.87  13.524
  58.179  12.672  74.043  12.069
#Mann= 3 , 0 , 0
       0    .035       0       0    .035       0  74.043    .035       0
Bank Sta=0,74.043
XS Rating Curve= 0
Exp/Cntr=.3,.1

Type RM Length L Ch R = 1 ,772     ,18,18,18
XS GIS Cut Line= 2
      1619716.63      4853269.05 1619674.4509079 4853356.9281085
#Sta/Elev= 24
       0  16.512   9.319  16.171  13.324  13.155  15.218  13.049  16.921  11.928
  18.263  11.368    23.3   11.15  24.776  11.089  28.218   9.896  30.717   9.706
  34.646    9.64  37.544   9.447   41.67   9.617  44.965   9.398  46.941   9.742
  48.119   9.814  50.887  11.391  52.311   11.41  57.323  11.476  61.564  13.475
  64.912  13.551  78.448  13.556  86.928  16.103  97.718  16.352
#Mann= 3 , 0 , 0
       0    .035       0       0    .035       0  97.718    .035       0
Bank Sta=0,97.718
XS Rating Curve= 0
Exp/Cntr=.3,.1

Type RM Length L Ch R = 3 ,771.5   ,,,
BEGIN DESCRIPTION:
Bretellina
END DESCRIPTION:
Bridge Culvert--1,0,-1,-1, 0
Deck Dist Width WeirC Skew NumUp NumDn MinLoCord MaxHiCord MaxSubmerge Is_Ogee
.5,17,1.44,0, 30, 30, , , .95, 0, 0,0,,
       0    9.31   13.32   13.32    15.2   16.91   18.21      24      24   24.74
   24.74   28.16   30.64   34.56   37.46   41.59   44.88   46.85   48.01    50.7
    50.7    51.5    51.5   57.16   61.39   64.72   78.24   78.24   86.69   97.47
   18.83   18.83   18.83   18.83   18.83   18.83   18.83   18.83   18.83   18.83
   18.83   18.83   18.83   18.83   18.83   18.83   18.83   18.83   18.83   18.83
   18.83   18.83   18.83   18.83   18.83   18.83   18.83   18.83   18.83   18.83
   16.51   16.17   13.15   15.28   15.28   15.28   15.28   15.28   11.07   11.08
   15.28   15.28   15.28   15.28   15.28   15.28   15.28   15.28   15.28   15.28
   11.42    11.4   15.28   15.28   15.28   15.28    15.2   13.56   15.28   15.28
       0    9.31   13.32   13.32    15.2   16.91   18.21      24      24   24.74
   24.74   28.16   30.64   34.56   37.46   41.59   44.88   46.85   48.01    50.7
    50.7    51.5    51.5   57.16   61.39   64.72   78.24   78.24   86.69   97.47
   18.83   18.83   18.83   18.83   18.83   18.83   18.83   18.83   18.83   18.83
   18.83   18.83   18.83   18.83   18.83   18.83   18.83   18.83   18.83   18.83
   18.83   18.83   18.83   18.83   18.83   18.83   18.83   18.83   18.83   18.83
   16.51   16.17   13.15   15.28   15.28   15.28   15.28   15.28   11.07   11.08
   15.28   15.28   15.28   15.28   15.28   15.28   15.28   15.28   15.28   15.28
   11.42    11.4   15.28   15.28   15.28   15.28    15.2   13.56   15.28   15.28
BR Coef=-1 , 0 , 0 ,1.25, 0 ,,,.8,-1,2,0,
WSPro=,,,, 1 ,,,, 0 ,,,, 0 ,,,,-1 ,-1 ,-1 , 0 , 0 , 0 , 0 , 0
BC Design=,, 0 ,, 0 ,,,,,,
BC HTab Sub Flow Pts= 40

Type RM Length L Ch R = 1 ,771.3   ,2.54,2.54,2.54
XS GIS Cut Line= 2
      1619716.63      4853269.05 1619674.4509079 4853356.9281085
#Sta/Elev= 24
       0  16.512   9.319  16.171  13.324  13.155  15.218  13.049  16.921  11.928
  18.263  11.368    23.3   11.15  24.776  11.089  28.218   9.896  30.717   9.706
  34.646    9.64  37.544   9.447   41.67   9.617  44.965   9.398  46.941   9.742
  48.119   9.814  50.887  11.391  52.311   11.41  57.323  11.476  61.564  13.475
  64.912  13.551  78.448  13.556  86.928  16.103  97.718  16.352
#Mann= 3 , 0 , 0
       0    .035       0       0    .035       0  97.718    .035       0
Bank Sta=0,97.718
XS Rating Curve= 0
Exp/Cntr=.3,.1

Type RM Length L Ch R = 1 ,771     ,23.45,23.45,23.45
XS GIS Cut Line= 2
      1619702.69      4853267.74 1619664.6481939  4853351.921868
#Sta/Elev= 30
       0  16.809   2.673  16.684   3.295  15.765   3.808  15.653   4.854  16.426
   7.585  14.818   8.864  13.762   9.888  13.412  16.185  12.938  18.025  11.678
  22.157  11.693  23.108   11.36  25.088  11.199  27.511  11.118  30.736  10.632
  32.827   9.645  36.491   9.597  40.067   9.523  44.125   9.523  49.012   9.394
  53.075   9.167  55.135    9.22  57.107   9.284  59.962  11.336  64.338  11.391
  68.553  13.363  74.098  13.456  78.106  15.767   87.48  16.392   94.64  16.308
#Mann= 3 , 0 , 0
       0    .035       0       0    .035       0   94.64    .035       0
Bank Sta=0,94.64
XS Rating Curve= 0
Exp/Cntr=.3,.1

Type RM Length L Ch R = 1 ,770     ,51.48,51.48,51.48
XS GIS Cut Line= 2
      1619639.99       4853284.8  1619679.968886 4853348.6082221
#Sta/Elev= 22
       0  12.654   8.578  12.797  11.429  14.058  17.537  14.246   25.28   11.15
   28.47  10.981  31.296   9.877   31.49   9.635  32.683   9.531  35.785   9.224
  38.915   9.513  42.032   9.422  45.351    9.58  46.888   9.607  49.062  11.175
  52.123  11.299  54.831  13.057   57.48  13.138  61.524   16.03  63.097  16.399
  70.268  16.359  75.438  16.167
#Mann= 3 , 0 , 0
       0    .035       0       0    .035       0  75.438    .035       0
Bank Sta=0,75.438
XS Rating Curve= 0
Exp/Cntr=.3,.1

Type RM Length L Ch R = 1 ,769     ,29.6,29.6,29.6
XS GIS Cut Line= 2
      1619595.76      4853332.04      1619662.08      4853383.67
#Sta/Elev= 27
       0  12.528   7.425  12.454  12.092  14.832  12.994  15.035  17.362  14.981
  18.593  14.693  25.049  11.408   29.93  10.878  31.218   10.03  31.339   9.752
  33.189   9.431  35.486   9.424  38.677   9.306  42.596    9.52  45.358   9.622
  46.861    9.63  48.397   9.697  50.997  10.892  55.455  11.391  58.554  13.033
  62.676  12.953  63.686  12.388  64.337  12.385  64.663  12.671  65.647   12.68
  71.839   16.36   84.23  16.265
#Mann= 3 , 0 , 0
       0    .035       0       0    .035       0   84.23    .035       0
Bank Sta=0,84.23
XS Rating Curve= 0
Exp/Cntr=.3,.1

Type RM Length L Ch R = 1 ,768     ,48.35,48.35,48.35
XS GIS Cut Line= 3
      1619582.12      4853358.11      1619649.12      4853410.25
 1619649.1278153 4853410.2560819
#Sta/Elev= 23
       0  12.378   7.106  12.334  12.624  12.269  22.699  12.355  23.192  10.535
  25.591    9.48  27.702   9.729  32.327   9.416  35.192   9.416  38.066   9.454
  40.165   9.728  42.878   9.743  45.445  10.867  49.632  11.276  53.289  12.957
  59.385  13.226  63.459  12.618  64.059  12.143  64.782  12.146  65.289  12.648
  66.384  12.755  72.637  16.483   85.36  16.418
#Mann= 3 , 0 , 0
       0    .035       0       0    .035       0   85.36    .035       0
Bank Sta=0,85.36
XS Rating Curve= 0
Exp/Cntr=.3,.1

Type RM Length L Ch R = 1 ,767     ,53.37,53.37,53.37
XS GIS Cut Line= 3
      1619551.63      4853395.97      1619610.63        4853445.
 1619610.6322297  4853445.001853
#Sta/Elev= 25
       0  12.622   6.339  12.891   8.821  14.882  12.394  14.843  19.633  11.164
  24.097  10.787  25.997  10.013  28.006   9.424  31.126   9.431  34.558   9.217
  37.674    9.23  40.265   9.272  41.485   9.739  43.096   9.823  45.202  10.941
  48.819  11.093  52.453  13.088  56.109  13.099  58.817  12.155  69.453  12.639
  73.433  12.502  74.119  12.004  74.666  12.018  75.154  12.517  76.953  12.678
#Mann= 3 , 0 , 0
       0    .035       0       0    .035       0  76.953    .035       0
Bank Sta=0,76.953
XS Rating Curve= 0
Exp/Cntr=.3,.1

Type RM Length L Ch R = 1 ,766     ,48.89,48.89,48.89
XS GIS Cut Line= 2
      1619515.06      4853434.32 1619572.5493112 4853482.7094203
#Sta/Elev= 21
       0  12.796   8.773  12.815  12.267  14.569  16.652  14.703  24.095  11.137
  27.677  10.978  30.472  10.032  30.783   9.742  32.587   9.237  35.419   9.229
  38.066    9.22  41.751   9.325   45.19    9.53  46.577   9.635  48.441  10.573
  52.961  11.009  57.001  13.156  60.733  13.158  62.678  12.319   69.07  12.267
  75.289  12.177
#Mann= 3 , 0 , 0
       0    .035       0       0    .035       0  75.289    .035       0
Bank Sta=0,75.289
XS Rating Curve= 0
Exp/Cntr=.3,.1

Type RM Length L Ch R = 1 ,765     ,84.19,84.19,84.19
XS GIS Cut Line= 2
      1619484.15       4853469.7 1619526.9092616 4853508.6993265
#Sta/Elev= 20
       0  12.569   3.995  12.602   7.846  14.496  12.211  14.496  19.983  11.141
  24.427  10.571  25.913  10.114   26.13    9.58  27.638   9.508  31.023   9.247
  34.433   9.165  36.342   9.118  39.084   9.374  41.344   9.635   42.53   9.515
  44.313  10.516  48.856  10.977  52.434  13.056  56.374  13.056  57.929  12.589
#Mann= 3 , 0 , 0
       0    .035       0       0    .035       0  57.929    .035       0
Bank Sta=0,57.929
XS Rating Curve= 0
Exp/Cntr=.3,.1

Type RM Length L Ch R = 1 ,764     ,19.92,19.92,19.92
XS GIS Cut Line= 3
      1619432.96      4853515.77 1619457.7043412 4853567.1917088
 1619463.8117765 4853579.8836918
#Sta/Elev= 24
       0  12.135   3.431  12.318   8.671  15.821  18.768  15.661  28.985  11.297
  32.445      11  35.963   9.901  36.197    9.47  37.579   9.523  40.922   9.318
  44.331   9.352  46.667    8.92  49.072   9.629   50.06   9.705  51.915   9.752
  56.661   9.925   59.22   9.965  59.295  12.896  62.404    12.9   62.59  10.164
  64.363  10.128  65.411  12.347  66.496  12.934  72.014  12.824
#Mann= 3 , 0 , 0
       0    .035       0       0    .035       0  72.014    .035       0
Bank Sta=0,72.014
XS Rating Curve= 0
Exp/Cntr=.3,.1

Type RM Length L Ch R = 1 ,763     ,56.61,56.61,56.61
XS GIS Cut Line= 2
       1619428.5      4853517.14 1619434.4296443 4853583.5160181
#Sta/Elev= 22
       0  11.993    2.76  12.077   8.267  15.686  18.487  15.889  28.491   11.29
  32.777  10.911   35.58  10.082  35.883   9.881  37.644   9.536  40.052   9.325
  42.756   9.224  44.848   8.925  46.351   9.245  49.841   9.707  55.699   9.819
  58.437   9.348  58.493  13.137  61.918  13.022  62.185  12.711  63.266  12.638
  63.398   9.934  67.426    9.95
#Mann= 3 , 0 , 0
       0    .035       0       0    .035       0  67.426    .035       0
Bank Sta=0,67.426
XS Rating Curve= 0
Exp/Cntr=.3,.1

Type RM Length L Ch R = 1 ,762     ,23.65,23.65,23.65
XS GIS Cut Line= 3
      1619379.36      4853532.17      1619374.24      4853594.51
 1619374.2397624 4853594.5128932
#Sta/Elev= 23
       0  10.323   5.322  10.316   5.571   12.17   6.306  12.228   6.473  13.117
   7.724  13.189   7.917   13.79   8.412  13.752   8.465   9.844   13.19   9.663
  15.555   9.449  16.974   9.524  20.247   9.527  24.193    9.27  27.282    9.12
  30.885   9.431  32.445   9.823   33.87  10.861  38.143  11.169  41.609   12.85
  46.031   12.98  47.731  12.597  62.963  12.069
#Mann= 3 , 0 , 0
       0    .035       0       0    .035       0  62.963    .035       0
Bank Sta=0,62.963
XS Rating Curve= 0
Exp/Cntr=.3,.1

Type RM Length L Ch R = 1 ,761     ,44.36,44.36,44.36
XS GIS Cut Line= 3
      1619352.68      4853536.12      1619359.95      4853604.25
  1619359.950531 4853604.2549766
#Sta/Elev= 18
       0  11.444   3.852  11.277   8.821  10.915  11.152   10.08  11.431   9.857
  13.089    9.63  15.834   9.424  18.592   8.925  22.614   9.323   24.79   9.531
  26.339   9.745  28.831   11.03  32.617  11.244  36.343  12.972  43.117  12.812
  44.466  12.068  60.335  11.789  68.955  11.791
#Mann= 3 , 0 , 0
       0    .035       0       0    .035       0  68.955    .035       0
Bank Sta=0,68.955
XS Rating Curve= 0
Exp/Cntr=.3,.1

Type RM Length L Ch R = 1 ,760     ,46.34,46.34,46.34
XS GIS Cut Line= 3
      1619297.78       4853549.2      1619339.63      4853620.24
 1619339.6300503 4853620.2400855
#Sta/Elev= 22
       0  13.092   1.723  14.056   9.426  13.867  13.996  11.344  18.866  10.903
  20.028  10.201   20.35   9.803  22.173   9.438  24.535   9.034  26.997   9.133
  29.942   9.431  32.089   9.535  34.318   9.745  35.615   9.818  37.877  10.956
  41.968  11.152   46.32  13.253  51.268  13.403  53.952   12.54  63.555  12.221
  73.696  12.138   83.34  12.102
#Mann= 3 , 0 , 0
       0    .035       0       0    .035       0   83.34    .035       0
Bank Sta=0,83.34
XS Rating Curve= 0
Exp/Cntr=.3,.1

Type RM Length L Ch R = 1 ,693     ,13.26,13.26,13.26
XS GIS Cut Line= 2
       1619259.1      4853568.11      1619290.24      4853629.23
#Sta/Elev= 18
       0   13.05 11.9201 14.1601 14.9599   13.51   18.69 11.6299 23.5799   11.12
   25.67 10.2599 26.1601  9.6201 28.3699  9.0901 32.6901  8.6999 38.5901    9.08
 41.1501    9.66    41.5 10.3501 42.3001    10.8 46.5201   11.12 50.7501    13.2
   56.05   13.46 57.9599 12.4099 68.6001 12.2301
#Mann= 3 , 0 , 0
       0    .035       0       0    .035       0 68.6001    .035       0
Bank Sta=0,68.6001
XS Rating Curve= 0
Exp/Cntr=.3,.1

Type RM Length L Ch R = 1 ,692     ,11.67,11.67,11.67
XS GIS Cut Line= 2
       1619254.6      4853571.62      1619269.72      4853637.12
#Sta/Elev= 17
       0 13.2999 10.6899 13.8401 15.5201    11.9 20.1799 11.2099 22.3799   10.29
   22.75  9.6701 24.3499    9.08 30.5099  8.6999   36.02    9.13 38.2801  9.6299
   38.78 10.0901 39.8099 10.7899 44.2301 11.1499 48.6001 13.3201 54.5299 13.1799
 56.4599 12.2901   67.22 12.1301
#Mann= 3 , 0 , 0
       0    .035       0       0    .035       0   67.22    .035       0
Bank Sta=0,67.22
XS Rating Curve= 0
Exp/Cntr=.3,.1
