HEC-RAS study ozz_def.prj: ozzeri

--- ozz_def.g02 (geometry) --- (continued)

Type RM Length L Ch R = 1 ,478     ,45.94,45.94,45.94
XS GIS Cut Line= 3
      1617417.25      4854355.94      1617397.08      4854419.71
 1617397.0796986 4854419.7109529
#Sta/Elev= 21
       0  12.069   8.649  12.145   12.66  10.255  17.305  10.295  23.366  10.639
  24.446  10.319  25.656   9.298  26.817   9.279   29.39    8.56  31.894   8.345
  33.758   8.179  35.536   8.345  37.544   8.999   38.68   9.323  40.327  10.438
  42.531  10.886  46.467  12.662  48.996  12.766  51.285  12.057  58.794   12.03
  67.061  12.013
#Mann= 3 , 0 , 0
       0    .035       0       0    .035       0  67.061    .035       0
Bank Sta=0,67.061
XS Rating Curve= 0
Exp/Cntr=.3,.1

Type RM Length L Ch R = 1 ,477     ,27.16,27.16,27.16
XS GIS Cut Line= 3
      1617373.64      4854343.08      1617358.66      4854394.26
 1617358.6588759 4854394.2638405
#Sta/Elev= 20
       0  12.546   6.245  12.766   7.611  12.638  12.632  10.239  16.911  10.434
   22.03  10.429  24.553   9.316  25.879    8.92  28.189   8.435  30.867   8.276
  33.615    8.53  35.397   8.481  38.092   9.075  39.194   9.964  42.901   10.23
  46.116  10.091   46.37  13.084  48.785  13.025  48.946  10.348  53.444  10.975
#Mann= 3 , 0 , 0
       0    .035       0       0    .035       0  53.444    .035       0
Bank Sta=0,53.444
XS Rating Curve= 0
Exp/Cntr=.3,.1

Type RM Length L Ch R = 1 ,476     ,50.35,50.35,50.35
XS GIS Cut Line= 3
      1617346.09      4854340.69      1617328.35      4854398.72
 1617328.3493866 4854398.7220064
#Sta/Elev= 21
       0  12.883   1.828  13.011   1.952    9.74   6.356   9.761  11.132   9.637
  13.521   9.857  15.055  10.022  15.907   9.557  17.692   9.383   19.83   8.668
  22.383   8.249  25.267   8.424  28.374   8.462  30.517   9.334  31.859   9.455
  35.273  11.293  38.617  11.813  39.694  12.431  43.826  12.366  53.173  11.947
  61.002  11.825
#Mann= 3 , 0 , 0
       0    .035       0       0    .035       0  61.002    .035       0
Bank Sta=0,61.002
XS Rating Curve= 0
Exp/Cntr=.3,.1

Type RM Length L Ch R = 1 ,475     ,66.68,66.68,66.68
XS GIS Cut Line= 3
       1617302.8      4854313.67      1617278.56       4854386.2
 1617278.5587642 4854386.2036976
#Sta/Elev= 25
       0  13.547   8.704  13.677   10.11  13.496   11.59  13.021  14.896  12.909
  18.126  11.253  20.973  10.927  23.975  10.339  26.195   9.744  27.044   9.499
  28.668   9.275  31.097   8.444  33.629   8.107  36.178   8.421  38.922   8.439
  40.621   9.247  42.034   9.401  44.066  10.289  46.553  11.307  51.782  11.808
  53.833  12.808  56.834  12.691  58.116  11.981  66.935  11.961  76.594  11.922
#Mann= 3 , 0 , 0
       0    .035       0       0    .035       0  76.594    .035       0
Bank Sta=0,76.594
XS Rating Curve= 0
Exp/Cntr=.3,.1

Type RM Length L Ch R = 1 ,474     ,51.6,51.6,51.6
XS GIS Cut Line= 2
      1617221.91      4854309.33 1617229.1895079 4854368.0160326
#Sta/Elev= 21
       0  12.212   8.284  12.627  10.488  12.482  12.284  12.374  17.261  10.802
   20.06   9.895   20.47   9.473   21.79   8.752  24.023   8.295  26.356   7.824
  29.386   8.371  31.563   8.958  34.736   9.281  36.749   9.424  39.641  10.064
  47.465  10.237  51.411  10.537  51.578  12.854  53.349  12.779  53.513      11
  59.386  11.682
#Mann= 3 , 0 , 0
       0    .035       0       0    .035       0  59.386    .035       0
Bank Sta=0,59.386
XS Rating Curve= 0
Exp/Cntr=.3,.1

Type RM Length L Ch R = 1 ,473.5   ,5.54,5.54,5.54
XS GIS Cut Line= 2
      1617168.21      4854326.38      1617186.27      4854384.01
#Sta/Elev= 23
       0   12.58    1.04 12.9799    7.78 12.7001  8.1601 12.4599   10.55   10.96
    13.2 10.6101 15.7999  9.4899 17.9299    9.13 19.0899    8.77 20.4499  8.4701
 21.9301  8.1799   23.22  8.3101 24.0399    8.46 26.8401  9.2501 28.0599    9.44
 29.6299    9.39   30.85  9.4601 32.1899  9.6701 37.6501 12.1899 43.0701 12.4901
 43.1499 12.4998   52.82 12.3599   60.55 12.1999
#Mann= 3 , 0 , 0
       0    .035       0  8.1601    .035       0 43.0701    .035       0
Bank Sta=8.1601,43.0701
XS Rating Curve= 0
Exp/Cntr=.3,.1

Type RM Length L Ch R = 1 ,473     ,8.15,8.15,8.15
XS GIS Cut Line= 2
      1617161.75       4854325.4      1617178.77      4854375.95
#Sta/Elev= 18
       0 13.4999  4.9399 13.6401 12.4998   13.89   12.53 13.8599 16.5701 10.6799
   18.84  9.9801 19.3801    9.44 21.2001  9.4601   23.18    9.45   24.69    9.45
   27.87    9.45 32.6499  9.2601   34.34     9.7 37.3401   10.85 41.1901 13.8099
   41.23 13.8501 47.8801   13.72 53.5701   13.47
#Mann= 3 , 0 , 0
       0    .035       0   12.53    .035       0 41.1901    .035       0
Bank Sta=12.53,41.1901
XS Rating Curve= 0
Exp/Cntr=.3,.1

Type RM Length L Ch R = 1 ,472.9   ,10,10,10
XS GIS Cut Line= 2
       1617151.6      4854314.11      1617179.34      4854391.64
#Sta/Elev= 18
       0 13.6599 12.8101 14.1101 15.8999 13.9199 19.8099   10.96   23.18    9.87
 23.5799    9.45 25.2201  9.2799 28.7201    8.87   31.11    8.77 34.9901  9.2699
 36.1499  9.4101 38.4901 10.4501   40.39 11.2499 44.0101 13.8099 44.2801 14.0101
   50.16 13.9001   57.82 13.5301   63.42   13.21
#Mann= 3 , 0 , 0
       0    .035       0       0    .035       0   63.42    .035       0
Bank Sta=0,63.42
XS Rating Curve= 0
Exp/Cntr=.3,.1

Type RM Length L Ch R = 3 ,472.8   ,,,
BEGIN DESCRIPTION:
ponte di meati
END DESCRIPTION:
Bridge Culvert--1,0,-1,-1, 0
Deck Dist Width WeirC Skew NumUp NumDn MinLoCord MaxHiCord MaxSubmerge Is_Ogee
.5,9,1.44,0, 11, 11, , , .95, 0, 0,0,,
       0 12.8101 15.8901   19.78   19.78      25   40.35   40.35 50.0899 57.7599
 63.3499
   14.36   14.36   14.36   14.36   14.36   14.36   14.36   14.36   14.36   14.36
   14.36
 12.5901 12.5901 12.5901   10.96 12.5901 12.5901 12.5901 11.2499 12.5901 12.5901
 12.5901
       0 12.8101 15.8901   19.78   19.78      25   40.35   40.35 50.0899 57.7599
 63.3499
   14.36   14.36   14.36   14.36   14.36   14.36   14.36   14.36   14.36   14.36
   14.36
 12.5901 12.5901 12.5901   10.96 12.5901 12.5901 12.5901 11.2499 12.5901 12.5901
 12.5901
BR Coef=-1 , 0 , 0 ,1.25, 0 ,,,.8,-1,2,0,
WSPro=,,,, 1 ,,,, 0 ,,,, 0 ,,,,-1 ,-1 ,-1 , 0 , 0 , 0 , 0 , 0
BC Design=,, 0 ,, 0 ,,,,,,
BC HTab Sub Flow Pts= 40

Type RM Length L Ch R = 1 ,472.7   ,15.54,15.54,15.54
XS GIS Cut Line= 2
       1617151.6      4854314.11      1617179.34      4854391.64
#Sta/Elev= 18
       0 13.6599 12.8101 14.1101 15.8999 13.9199 19.8099   10.96   23.18    9.87
 23.5799    9.45 25.2201  9.2799 28.7201    8.87   31.11    8.77 34.9901  9.2699
 36.1499  9.4101 38.4901 10.4501   40.39 11.2499 44.0101 13.8099 44.2801 14.0101
   50.16 13.9001   57.82 13.5301   63.42   13.21
#Mann= 3 , 0 , 0
       0    .035       0       0    .035       0   63.42    .035       0
Bank Sta=0,63.42
XS Rating Curve= 0
Exp/Cntr=.3,.1

Type RM Length L Ch R = 1 ,472     ,52.56,52.56,52.56
XS GIS Cut Line= 2
      1617131.94      4854313.08      1617151.69      4854396.57
#Sta/Elev= 20
       0  13.319  11.459  13.357  19.657  13.216   25.99  11.623  31.135  10.951
  35.277   9.759  35.511   9.646  38.073    9.28  41.947   8.475  44.047   8.879
  46.807    8.07   48.79   8.376  51.218   9.512  54.796  10.007  56.697  10.699
  62.703  10.636   68.74  10.659  73.733  11.908  78.561  12.296   85.86  12.419
#Mann= 3 , 0 , 0
       0    .035       0       0    .035       0   85.86    .035       0
Bank Sta=0,85.86
XS Rating Curve= 0
Exp/Cntr=.3,.1

Type RM Length L Ch R = 1 ,471     ,49.97,49.97,49.97
XS GIS Cut Line= 2
      1617082.32      4854339.62 1617104.5590596 4854407.1371449
#Sta/Elev= 21
       0   12.28   8.336  12.528   9.722  13.096   13.87  12.897  16.719  11.304
  20.718  10.833  22.764   9.611  24.723   9.278  28.013    8.38  31.224   7.879
  33.104   8.475  36.048   9.277  38.739   9.662  40.912  10.429  45.461  10.461
  51.764  10.447  58.207  10.682  61.939  10.845  65.158  10.895  67.265  10.861
  71.297  10.884
#Mann= 3 , 0 , 0
       0    .035       0       0    .035       0  71.297    .035       0
Bank Sta=0,71.297
XS Rating Curve= 0
Exp/Cntr=.3,.1

Type RM Length L Ch R = 1 ,470     ,37.63,37.63,37.63
XS GIS Cut Line= 2
      1617036.92      4854355.84 1617052.5190528  4854421.486014
#Sta/Elev= 16
       0  10.325   6.823  10.241  12.622  10.136  18.103   9.543  20.017   8.978
  23.259    8.74  26.671   8.427  29.063   8.439  30.687   8.854  33.455   8.904
  35.621  10.323  41.743  10.257  48.418  10.299  52.326  10.537  57.893   12.16
  67.496  12.332
#Mann= 3 , 0 , 0
       0    .035       0       0    .035       0  67.496    .035       0
Bank Sta=0,67.496
XS Rating Curve= 0
Exp/Cntr=.3,.1

Type RM Length L Ch R = 6 ,469.55  ,,,
Lateral Weir Pos= 3
Lateral Weir End=                ,                ,        ,c01
Lateral Weir Distance=1
Lateral Weir WD=3.0001
Lateral Weir Coef=1.66
Lateral Weir Is Ogee= 0
Lateral Weir WSCriteria=-1
Lateral Weir SE= 6
       0 15.0001       1 15.0001       1 11.5001     101 11.5001     101 15.0001
102.0001 15.0001

Type RM Length L Ch R = 1 ,469     ,68.65,68.65,68.65
XS GIS Cut Line= 2
       1616999.1      4854348.32 1617014.2692476 4854427.6360659
#Sta/Elev= 17
       0  11.783  16.072  11.661   23.73  11.361  27.933  10.857  36.038  10.383
  36.392   9.574  39.235   8.832  43.338   8.455  47.215   8.815  49.648   8.984
  51.784   9.341  52.922  10.324  58.119  10.315  62.123  10.255  65.564  10.908
  69.069  11.963  80.796  12.279
#Mann= 3 , 0 , 0
       0    .035       0       0    .035       0  80.796    .035       0
Bank Sta=0,80.796
XS Rating Curve= 0
Exp/Cntr=.3,.1

Type RM Length L Ch R = 6 ,468.55  ,,,
Lateral Weir Pos= 0
Lateral Weir End=                ,                ,        ,c02
Lateral Weir Distance=1
Lateral Weir WD=3.0001
Lateral Weir Coef=1.66
Lateral Weir Is Ogee= 0
Lateral Weir WSCriteria=-1
Lateral Weir SE= 6
       0 15.0001       1 15.0001       1 12.4998301.0001 12.4998301.0001 15.0001
302.0001 15.0001

Type RM Length L Ch R = 1 ,468     ,26.77,26.77,26.77
XS GIS Cut Line= 3
      1616930.16      4854367.99      1616947.38      4854434.63
 1616947.3807501  4854434.632903
#Sta/Elev= 22
       0  12.471  20.049  12.454  22.897  12.646  27.346   10.41   33.38  10.583
  34.441  10.164  34.849   9.322  36.659   8.518  39.669   8.745   41.92   8.486
  44.884   8.427   47.26   8.805  49.406   9.137  49.989   9.847  51.958   10.23
  55.209  10.394  57.344  10.583  59.921  11.242   61.87  12.824  63.073  12.829
  65.182  12.035  68.943  12.054
#Mann= 3 , 0 , 0
       0    .035       0       0    .035       0  68.943    .035       0
Bank Sta=0,68.943
XS Rating Curve= 0
Exp/Cntr=.3,.1

Type RM Length L Ch R = 1 ,467     ,25.46,25.46,25.46
XS GIS Cut Line= 3
      1616909.08      4854386.31      1616919.11      4854437.84
  1616919.110172 4854437.8408837
#Sta/Elev= 19
       0  12.229   6.088  11.275  12.404  10.697  21.564  10.514  23.075   9.896
  23.488   9.424  24.919   9.272  27.325   8.298  29.292   8.798  31.337   8.336
    33.3   8.279  35.333   8.444  37.166   9.072  38.421   9.996  42.205  10.394
  46.322  10.903  49.873  13.034   51.27  12.944  52.581  12.522
#Mann= 3 , 0 , 0
       0    .035       0       0    .035       0  52.581    .035       0
Bank Sta=0,52.581
XS Rating Curve= 0
Exp/Cntr=.3,.1

Type RM Length L Ch R = 1 ,466     ,41.11,41.11,41.11
XS GIS Cut Line= 2
      1616884.09      4854388.75 1616901.7497276 4854464.3588336
#Sta/Elev= 18
       0  10.598    14.5   10.27  17.331   10.08  26.849   9.466  29.501    8.96
  31.395   8.184  33.426   8.077  35.417   8.126  37.408   8.185  39.197   9.024
  41.107   9.241  42.649   9.995  46.755  10.208  49.643  10.303  54.312  12.833
  56.716  12.951  58.784  12.136  77.999  12.144
#Mann= 3 , 0 , 0
       0    .035       0       0    .035       0  77.999    .035       0
Bank Sta=0,77.999
XS Rating Curve= 0
Exp/Cntr=.3,.1

Type RM Length L Ch R = 1 ,465     ,66.09,66.09,66.09
XS GIS Cut Line= 2
      1616840.47       4854406.8 1616863.7596367 4854467.0190607
#Sta/Elev= 20
       0  12.309  10.368  12.286  12.176   12.18  16.552  10.478  22.126   10.46
  22.844  10.248  23.167   9.486  25.079   8.382  27.351   7.959  29.426   7.955
  32.404   8.206  34.239   9.322  36.736   9.365  38.571    9.98  43.709  10.059
   47.26  10.236  50.768  10.196  53.299  10.635  58.029  10.806  64.659  10.867
#Mann= 3 , 0 , 0
       0    .035       0       0    .035       0  64.659    .035       0
Bank Sta=0,64.659
XS Rating Curve= 0
Exp/Cntr=.3,.1

Type RM Length L Ch R = 1 ,464     ,58.21,58.21,58.21
XS GIS Cut Line= 3
      1616772.81      4854417.35      1616807.99       4854505.6
 1616807.9900367 4854505.6000921
#Sta/Elev= 22
       0  12.025  17.293  12.342  25.732  12.437   27.02  12.302  32.079  10.568
  39.161  10.145  40.193   9.889  40.696   9.452  42.295   8.671  44.652   8.079
  46.729   8.062  48.673   8.097  50.734   8.132   52.09   8.754  54.191   9.289
  56.128   10.25  60.636  10.093  66.205  12.841  68.068   12.86  70.197  12.267
  74.015  12.259   95.03  12.182
#Mann= 3 , 0 , 0
       0    .035       0       0    .035       0   95.03    .035       0
Bank Sta=0,95.03
XS Rating Curve= 0
Exp/Cntr=.3,.1

Type RM Length L Ch R = 1 ,463     ,56.84,56.84,56.84
XS GIS Cut Line= 3
      1616719.01      4854441.33      1616747.09      4854512.36
 1616747.0906984 4854512.3617667
#Sta/Elev= 22
       0  12.304  17.504  12.513  24.519  12.342  29.879  10.323  33.402  10.187
  37.709   10.32  39.201   9.436  40.975   9.096  43.548   8.149  46.475   7.986
  48.517   7.925  50.944   8.306  52.618   8.829  53.676    9.76  57.176  10.125
  60.708   10.12   63.29  10.666  63.653  12.824  66.202   12.73  66.302   10.77
  71.333  11.212  76.532  11.383
#Mann= 3 , 0 , 0
       0    .035       0       0    .035       0  76.532    .035       0
Bank Sta=0,76.532
XS Rating Curve= 0
Exp/Cntr=.3,.1

Type RM Length L Ch R = 1 ,462     ,50.05,50.05,50.05
XS GIS Cut Line= 2
      1616666.82      4854465.44 1616698.3499608 4854538.8199089
#Sta/Elev= 24
       0  12.022  16.845  12.174  18.887  13.133  20.117  13.018  21.483  12.629
  26.057  10.215  34.051  10.129  34.694  10.404  36.153  10.008  36.405   9.332
  38.313   8.798  40.777   8.364  43.666   7.774  45.673   7.916  47.709   8.294
  48.667   9.057  49.728   9.117  50.385   9.902  55.391  10.326  60.512  12.923
  62.286   12.85  64.497  12.241  70.564  12.132   79.93  12.168
#Mann= 3 , 0 , 0
       0    .035       0       0    .035       0   79.93    .035       0
Bank Sta=0,79.93
XS Rating Curve= 0
Exp/Cntr=.3,.1

Type RM Length L Ch R = 1 ,461     ,32.54,32.54,32.54
XS GIS Cut Line= 2
      1616626.76       4854495.1 1616653.9688562 4854563.5771214
#Sta/Elev= 23
       0  12.102   6.571  11.547   8.615  10.803   9.788  11.797  11.848  12.128
  12.619    10.6  14.952  10.156  23.946   9.882  24.504   9.329  26.546   8.535
  28.212   8.152  31.194   8.103   33.21    8.14  35.242   8.371  36.823    9.02
  38.035   9.196   38.91   9.733  45.727  10.242  50.234  12.908    51.3  12.925
  52.872  12.606  60.318   12.48  74.067  12.288
#Mann= 3 , 0 , 0
       0    .035       0       0    .035       0  74.067    .035       0
Bank Sta=0,74.067
XS Rating Curve= 0
Exp/Cntr=.3,.1

Type RM Length L Ch R = 1 ,460     ,65.78,65.78,65.78
XS GIS Cut Line= 3
       1616589.2      4854504.09      1616621.65      4854566.34
  1616621.650462 4854566.3408863
#Sta/Elev= 21
       0  12.125  15.969  12.353  16.951  12.869  20.379   12.78  24.233  10.475
   30.66  10.269  31.621   9.531  33.828     8.6  36.014   8.169  38.105   8.059
  40.073   8.152  42.175   8.539  44.328   9.088  46.493   9.322  47.736   9.882
  54.629  10.087   59.05  10.695  59.276  12.967  61.055  12.942  61.113  11.059
  70.571  11.248
#Mann= 3 , 0 , 0
       0    .035       0       0    .035       0  70.571    .035       0
Bank Sta=0,70.571
XS Rating Curve= 0
Exp/Cntr=.3,.1

Type RM Length L Ch R = 6 ,459.55  ,,,
Lateral Weir Pos= 0
Lateral Weir End=                ,                ,        ,c02
Lateral Weir Distance=1
Lateral Weir WD=3.0001
Lateral Weir Coef=1.66
Lateral Weir Is Ogee= 0
Lateral Weir WSCriteria=-1
Lateral Weir SE= 6
       0 15.0001       1 15.0001       1 12.9001      51 12.9001      51 15.0001
 52.0001 15.0001

Type RM Length L Ch R = 1 ,459     ,40.5,40.5,40.5
XS GIS Cut Line= 2
      1616539.58      4854542.91 1616564.3088607 4854603.1072266
#Sta/Elev= 23
       0  12.184   3.556   11.04   5.719  10.581    6.19  12.323    6.36  10.602
   9.422  10.419   9.711  10.373  16.726  10.358  20.394  10.186  22.011   9.774
  22.236   9.379  24.139   9.104  26.777   8.374  28.805   7.924  30.778   8.251
  31.651   8.328   34.66   8.965  35.393   9.691  37.781  10.141  43.048  10.246
  47.826   12.74  54.179  13.016  65.817  12.949
#Mann= 3 , 0 , 0
       0    .035       0       0    .035       0  65.817    .035       0
Bank Sta=0,65.817
XS Rating Curve= 0
Exp/Cntr=.3,.1

Type RM Length L Ch R = 1 ,458     ,45.74,45.74,45.74
XS GIS Cut Line= 2
      1616504.76        4854572. 1616536.4179647 4854627.3764399
#Sta/Elev= 16
       0  10.852   2.833  10.446  10.964  10.303  13.006   9.497  15.503   8.849
  18.823   8.199  21.887   8.368  24.112   8.589  25.829   8.756  26.863   8.991
  28.858  10.361  36.648  10.987  40.193  12.841   41.96  13.152  54.087  13.024
  63.896  13.039
#Mann= 3 , 0 , 0
       0    .035       0       0    .035       0  63.896    .035       0
Bank Sta=0,63.896
XS Rating Curve= 0
Exp/Cntr=.3,.1

Type RM Length L Ch R = 1 ,457     ,33.2,33.2,33.2
XS GIS Cut Line= 2
      1616453.66      4854579.44 1616492.1089352 4854636.2484268
#Sta/Elev= 21
       0  13.014  12.449  13.046  23.328  12.586  27.556  10.262  34.431  10.289
  35.107    9.62  36.875   8.341  39.263   7.917  41.264   7.738  43.199   7.698
  45.929   8.853  47.507   9.268  48.598   9.022   49.83   9.943  53.128  10.114
  59.706  10.201  61.106  10.743  61.305  13.097  63.163  13.039  63.327  11.376
  68.658   11.97
#Mann= 3 , 0 , 0
       0    .035       0       0    .035       0  68.658    .035       0
Bank Sta=0,68.658
XS Rating Curve= 0
Exp/Cntr=.3,.1

Type RM Length L Ch R = 1 ,456     ,41.98,41.98,41.98
XS GIS Cut Line= 3
      1616436.59      4854616.37       1616468.7      4854666.28
 1616468.7000557 4854666.2800866
#Sta/Elev= 18
       0  11.484   3.155  11.025   6.045  10.577  13.238  10.136   13.83    9.29
  15.826    8.82  18.124   8.142  20.126   7.987  23.175    8.02   25.57   8.313
  27.085   8.946  28.797   9.689   30.93  10.331  35.586  10.351  40.847  12.876
  44.229  13.235  54.168  13.269   60.06  13.226
#Mann= 3 , 0 , 0
       0    .035       0       0    .035       0   60.06    .035       0
Bank Sta=0,60.06
XS Rating Curve= 0
Exp/Cntr=.3,.1

Type RM Length L Ch R = 1 ,455     ,79.96,79.96,79.96
XS GIS Cut Line= 3
      1616400.42      4854640.62      1616442.73      4854689.92
 1616442.7312372 4854689.9214416
#Sta/Elev= 17
       0  10.581   3.378  10.396   6.322     9.8   8.785   9.766  13.763   9.842
  15.646   9.482  18.026   9.024  19.968   8.207  22.958   8.143  24.978   8.185
  27.571   8.745  29.042   9.028  30.626  10.224  38.741   10.45   43.48   13.03
  50.869  13.155  65.202  13.028
#Mann= 3 , 0 , 0
       0    .035       0       0    .035       0  65.202    .035       0
Bank Sta=0,65.202
XS Rating Curve= 0
Exp/Cntr=.3,.1

Type RM Length L Ch R = 1 ,454     ,60.57,60.57,60.57
XS GIS Cut Line= 2
      1616333.75      4854666.77  1616361.228331 4854724.7764767
#Sta/Elev= 20
       0  14.241  15.387  14.394  17.506  13.117  21.896  12.989  25.002  11.014
  33.478  10.762  35.721  10.146  37.086   9.415  40.065   9.157   42.04   8.656
  44.059   8.165  46.124   8.137  48.148   7.913   50.56   8.597  52.012   9.155
  53.359  10.171  57.905  10.564  61.319  12.713  62.454  12.923  64.286  12.914
#Mann= 3 , 0 , 0
       0    .035       0       0    .035       0  64.286    .035       0
Bank Sta=0,64.286
XS Rating Curve= 0
Exp/Cntr=.3,.1

Type RM Length L Ch R = 6 ,453.55  ,,,
Lateral Weir Pos= 3
Lateral Weir End=                ,                ,        ,c01
Lateral Weir Distance=1
Lateral Weir WD=3.0001
Lateral Weir Coef=1.66
Lateral Weir Is Ogee= 0
Lateral Weir WSCriteria=-1
Lateral Weir SE= 6
       0 15.0001       1 15.0001       1 12.7001     101 12.7001     101 15.0001
102.0001 15.0001

Type RM Length L Ch R = 1 ,453     ,48.74,48.74,48.74
XS GIS Cut Line= 2
       1616285.6      4854682.38 1616297.5792384 4854744.1060754
#Sta/Elev= 29
       0  13.119   3.251  12.423   4.274   12.31   7.264  13.647    9.93   15.24
  11.098  15.275  14.183  13.284  18.879  13.105   21.49    11.2  30.208  10.653
  34.284   9.543  37.526    9.37  39.819   8.455  41.756   7.836  43.802    7.76
  45.866   7.932  47.467   8.363  49.045   9.037  49.551  10.025  50.887  10.434
  55.497  10.833  58.192  12.486   59.34  12.905  60.607  13.115  62.462  13.959
  62.535  14.608   62.78  14.606  62.819  14.821  63.416  14.928
#Mann= 3 , 0 , 0
       0    .035       0       0    .035       0  63.416    .035       0
Bank Sta=0,63.416
XS Rating Curve= 0
Exp/Cntr=.3,.1

Type RM Length L Ch R = 1 ,452     ,2.21,2.21,2.21
XS GIS Cut Line= 2
      1616236.27      4854701.75 1616254.8992227 4854745.8881584
#Sta/Elev= 22
       0  12.358   2.502  12.191    5.64  11.053  12.372  10.986  12.868  13.922
  13.077  13.929  13.173  13.246  14.642  13.227  14.842  13.932  15.077   13.94
  15.425    10.3  17.116   9.677  23.075   9.376  24.997   8.572  27.601   8.348
  30.594   8.679  32.618    8.65  35.414   9.278  36.457   9.313   37.23   9.993
   42.03  10.168  49.268  10.292
#Mann= 3 , 0 , 0
       0    .035       0       0    .035       0  49.268    .035       0
Bank Sta=0,49.268
XS Rating Curve= 0
Exp/Cntr=.3,.1

Type RM Length L Ch R = 1 ,451     ,4.8,4.8,4.8
XS GIS Cut Line= 2
      1616214.72      4854721.49 1616300.7404245 4854744.1774745
#Sta/Elev= 21
       0  12.483  11.775   11.28  21.446    9.92  21.689   9.453  24.572   8.399
  27.419   8.454  29.438   8.338  31.464   8.474  33.476   8.731  35.457   8.762
  39.068   9.062  40.843   9.958  46.599  10.469  52.652  10.493  60.869  10.399
  71.538  10.788  79.951  12.698   83.78  13.059   85.48  13.808   85.54  14.666
   89.06  14.637
#Mann= 3 , 0 , 0
       0    .035       0       0    .035       0   89.06    .035       0
Bank Sta=0,89.06
XS Rating Curve= 0
Exp/Cntr=.3,.1

Type RM Length L Ch R = 1 ,450.2   ,20,20,20
XS GIS Cut Line= 3
      1616209.08      4854743.91      1616255.47      4854756.57
 1616255.4737611 4854756.5710264
#Sta/Elev= 17
       0  12.314  1.9897  12.414  2.5733  13.487  4.2354  11.404  11.872  10.222
  15.245  9.3639   17.02  8.9569  18.792  8.8459  21.127  8.9739  23.657  9.0299
  25.828  9.1179  28.164   9.154  32.607  9.6339  38.394  10.558  44.824  11.089
  48.134  12.956  48.134   13.96
#Mann= 3 , 0 , 0
       0    .035       0       0    .035       0  48.134    .035       0
Bank Sta=0,48.134
XS Rating Curve= 0
Exp/Cntr=.3,.1

Type RM Length L Ch R = 3 ,450.1   ,,,
BEGIN DESCRIPTION:
A11
END DESCRIPTION:
Bridge Culvert--1,0,-1,-1, 0
Deck Dist Width WeirC Skew NumUp NumDn MinLoCord MaxHiCord MaxSubmerge Is_Ogee
.5,19,1.44,0, 27, 27, , , .95, 0, 0,0,,
       0   11.77   14.25   14.25   15.25   15.25   21.44   21.65   24.52   27.36
   29.38   32.61   32.61   33.61   33.61   35.39      39   40.77   46.53   52.58
    60.8   71.46   79.87   83.69   85.39   85.44   88.97
   14.63   14.63   14.63   14.63   14.63   14.63   14.63   14.63   14.63   14.63
   14.63   14.63   14.63   14.63   14.63   14.63   14.63   14.63   14.63   14.63
   14.63   14.63   14.63   14.63   14.63   14.63   14.63
   13.96   13.96   13.96     9.4    9.36   13.96   13.96   13.96   13.96   13.96
   13.96   13.96    9.63     9.7   13.96   13.96   13.96   13.96   13.96   13.96
   13.96   13.96   13.96   13.96   13.96   13.96   13.96
       0   11.77   14.25   14.25   15.25   15.25   21.44   21.65   24.52   27.36
   29.38   32.61   32.61   33.61   33.61   35.39      39   40.77   46.53   52.58
    60.8   71.46   79.87   83.69   85.39   85.44   88.97
   14.63   14.63   14.63   14.63   14.63   14.63   14.63   14.63   14.63   14.63
   14.63   14.63   14.63   14.63   14.63   14.63   14.63   14.63   14.63   14.63
   14.63   14.63   14.63   14.63   14.63   14.63   14.63
   13.96   13.96   13.96     9.4    9.36   13.96   13.96   13.96   13.96   13.96
   13.96   13.96    9.63     9.7   13.96   13.96   13.96   13.96   13.96   13.96
   13.96   13.96   13.96   13.96   13.96   13.96   13.96
BR Coef=-1 , 0 , 0 ,1.25, 0 ,,,.8,-1,2,0,
WSPro=,,,, 1 ,,,, 0 ,,,, 0 ,,,,-1 ,-1 ,-1 , 0 , 0 , 0 , 0 , 0
BC Design=,, 0 ,, 0 ,,,,,,
BC HTab Sub Flow Pts= 40

Type RM Length L Ch R = 1 ,450     ,1.6,1.6,1.6
XS GIS Cut Line= 2
      1616209.08      4854743.91      1616255.47      4854756.57
#Sta/Elev= 16
       0   12.31    1.99 12.4099  2.5701 13.4901  4.2401 11.4001 11.8701 10.2199
   15.24  9.3601   17.02  8.9599   18.79  8.8499   21.13    8.97 23.6601    9.03
   25.83  9.1199 28.1599  9.1501 32.6099  9.6299 38.3899 10.5601 44.8199 11.0901
 48.1301 12.9601
#Mann= 3 , 0 , 0
       0    .035       0       0    .035       0 48.1301    .035       0
Bank Sta=0,48.1301
XS Rating Curve= 0
Exp/Cntr=.3,.1

Type RM Length L Ch R = 1 ,449     ,12.65,12.65,12.65
XS GIS Cut Line= 2
      1616252.01      4854761.65 1616210.9346107 4854746.8216645
#Sta/Elev= 14
       0  10.161   4.929  10.083   8.529    9.97  15.487   9.775  18.999   8.983
  20.799   8.847  22.879   9.835  24.261   9.601  25.017   8.934  27.876   8.886
  32.376   9.302  34.786  10.542  41.696  10.773  44.135  12.692
#Mann= 3 , 0 , 0
       0    .035       0       0    .035       0  44.135    .035       0
Bank Sta=0,44.135
XS Rating Curve= 0
Exp/Cntr=.3,.1

Type RM Length L Ch R = 1 ,448     ,1.26,1.26,1.26
XS GIS Cut Line= 2
      1616207.54      4854757.42 1616188.1418399 4854750.8567127
#Sta/Elev= 14
       0  12.692   2.439  10.773   9.348  10.542  11.758   9.302  16.259   8.888
  19.117   8.934  19.874   9.601  21.256   9.835  23.335   8.848  25.135   8.983
  28.648   9.776  35.606    9.97  39.206  10.083  44.135  10.161
#Mann= 3 , 0 , 0
       0    .035       0       0    .035       0  44.135    .035       0
Bank Sta=0,44.135
XS Rating Curve= 0
Exp/Cntr=.3,.1

Type RM Length L Ch R = 1 ,447.8   ,7,7,7
#Sta/Elev= 20
       0  13.768     .48  13.563    4.16  10.685    5.05   9.985    8.95   9.982
    9.92   9.434   11.53   8.936   13.89   8.894   14.83   9.034   18.86   9.062
   22.63   8.867   24.32   9.003   26.07   8.709   27.74   9.325   28.15   9.784
   32.25   9.986   33.16  10.694   36.88  13.639   40.84   14.09   45.15  14.166
#Mann= 3 , 0 , 0
       0    .035       0       0    .035       0   45.15    .035       0
Bank Sta=0,45.15
XS Rating Curve= 0
Exp/Cntr=.3,.1

Type RM Length L Ch R = 3 ,447.6   ,,,
BEGIN DESCRIPTION:
Ponte FFSS
END DESCRIPTION:
Bridge Culvert--1,0,-1,-1, 0
Deck Dist Width WeirC Skew NumUp NumDn MinLoCord MaxHiCord MaxSubmerge Is_Ogee
.5,6,1.44,0, 30, 30, , , .95, 0, 0,0,,
       0     .48    4.16    5.05    5.05    6.36    8.12    9.15   10.79   12.85
   12.85   13.89   15.01   15.01   16.91   18.01   21.15   23.15   23.15   24.84
   24.84   26.75   28.72   30.75   32.65   32.65   33.15   36.87   40.84   45.15
   14.17   14.17   14.17   14.17   14.17   14.17   14.17   14.17   14.17   14.17
   14.17   14.17   14.17   14.17   14.17   14.17   14.17   14.17   14.17   14.17
   14.17   14.17   14.17   14.17   14.17   14.17   14.17   14.17   14.17   14.17
   13.77   13.56   10.69    9.98   11.12   11.85   12.53   12.66   12.39   11.12
     8.9    8.89    9.03   11.17   12.28   12.71   12.32   11.14     8.9       9
    11.2   12.39   12.76   12.45   11.12   10.65   10.69   13.64   14.09    14.1
       0     .48    4.16    5.05    5.05    6.36    8.12    9.15   10.79   12.85
   12.85   13.89   15.01   15.01   16.91   18.01   21.15   23.15   23.15   24.84
   24.84   26.75   28.72   30.75   32.65   32.65   33.15   36.87   40.84   45.15
   14.17   14.17   14.17   14.17   14.17   14.17   14.17   14.17   14.17   14.17
   14.17   14.17   14.17   14.17   14.17   14.17   14.17   14.17   14.17   14.17
   14.17   14.17   14.17   14.17   14.17   14.17   14.17   14.17   14.17   14.17
   13.77   13.56   10.69    9.98   11.12   11.85   12.53   12.66   12.39   11.12
     8.9    8.89    9.03   11.17   12.28   12.71   12.32   11.14     8.9       9
    11.2   12.39   12.76   12.45   11.12   10.65   10.69   13.64   14.09    14.1
BR Coef=-1 , 0 , 0 ,1.25, 0 ,,,.8,-1,2,0,
WSPro=,,,, 1 ,,,, 0 ,,,, 0 ,,,,-1 ,-1 ,-1 , 0 , 0 , 0 , 0 , 0
BC Design=,, 0 ,, 0 ,,,,,,

Type RM Length L Ch R = 1 ,447.5   ,1,1,1
#Sta/Elev= 20
       0   13.77     .48   13.56    4.16   10.69    5.05    9.98    8.95    9.98
    9.91    9.43   11.53    8.94   13.89    8.89   14.83    9.03   18.86    9.06
   22.63    8.87   24.32       9   26.07    8.71   27.74    9.32   28.15    9.78
   32.25    9.99   33.15   10.69   36.87   13.64   40.84   14.09   45.15   14.17
#Mann= 3 , 0 , 0
       0    .035       0       0    .035       0   45.15    .035       0
Bank Sta=0,45.15
XS Rating Curve= 0
Exp/Cntr=.3,.1

Type RM Length L Ch R = 1 ,447     ,22.52,22.52,22.52
XS GIS Cut Line= 2
      1616197.96      4854765.35   1616243.41606 4854778.4688629
#Sta/Elev= 23
       0   13.93   7.301  13.652  11.424  10.153   11.97   9.828  13.246   9.693
  14.164   9.302  17.427   9.098  19.939   9.261  20.926   9.185   21.91   9.018
  24.736   8.924  27.007   8.955  29.792   8.961  30.821   9.092  31.763   9.052
  33.575    9.09  35.883   8.981  37.122   9.445  37.754   9.904  39.675  10.194
  40.519  10.543   44.32  13.885  48.346  13.991
#Mann= 3 , 0 , 0
       0    .035       0       0    .035       0  48.346    .035       0
Bank Sta=0,48.346
XS Rating Curve= 0
Exp/Cntr=.3,.1

Type RM Length L Ch R = 1 ,446     ,54.71,54.71,54.71
XS GIS Cut Line= 2
      1616187.05      4854782.53 1616236.6142526  4854800.147957
#Sta/Elev= 16
       0  14.116  10.574  13.245  16.939  10.836  19.015   9.497  20.785   8.871
  23.585   8.676   27.33   8.542  30.208    8.63  32.921   8.129  36.218   8.856
  36.928   8.978  38.704  10.103  41.168  10.505  50.619  10.771  50.707  13.454
  52.724  13.479
#Mann= 3 , 0 , 0
       0    .035       0       0    .035       0  52.724    .035       0
Bank Sta=0,52.724
XS Rating Curve= 0
Exp/Cntr=.3,.1

Type RM Length L Ch R = 1 ,398     ,49.84,49.84,49.84
XS GIS Cut Line= 2
      1616157.98      4854821.61 1616208.1291475 4854852.2994783
#Sta/Elev= 22
       0  13.158   2.047  13.225    2.67  13.625  14.493  13.649  15.346  13.417
  17.999  13.085  21.263  11.008    26.1  11.015  29.094   9.393   29.49   8.993
  33.091   8.367  34.309     8.3  36.477   8.195  38.486   8.206  40.501   8.173
  42.534   8.367  44.547   8.984  45.875    8.89   47.87  10.143  52.695  10.379
  58.469  13.373  60.119  13.565
#Mann= 3 , 0 , 0
       0    .035       0       0    .035       0  60.119    .035       0
Bank Sta=0,60.119
XS Rating Curve= 0
Exp/Cntr=.3,.1

Type RM Length L Ch R = 1 ,397     ,52.53,52.53,52.53
XS GIS Cut Line= 2
      1616126.49      4854852.05 1616177.6984868 4854896.2486939
#Sta/Elev= 22
       0    12.9  17.274  13.182  17.384  13.291  21.184   13.22  24.498  11.128
  29.751  10.774  34.576   9.211  34.863   9.009  36.813   9.104  37.956   8.902
  39.822   8.524  40.036   7.986  42.295   7.873  44.299   8.079   46.51   8.374
  47.753   8.953  48.961   8.838  49.611   9.774  55.102  10.213  59.912  12.629
  63.259  12.833  67.688  12.925
#Mann= 3 , 0 , 0
       0    .035       0       0    .035       0  67.688    .035       0
Bank Sta=0,67.688
XS Rating Curve= 0
Exp/Cntr=.3,.1

Type RM Length L Ch R = 1 ,396     ,57.63,57.63,57.63
XS GIS Cut Line= 2
      1616096.41      4854876.71      1616129.67      4854929.81
#Sta/Elev= 24
       0  12.742  15.078  12.652  15.335  12.373  15.753  12.233  17.913  12.742
  19.674  12.515  21.572  11.842  25.076  11.638  26.708  11.223  31.296   9.419
  33.602   9.152    36.3   9.072  37.723   8.966  38.869   8.234  41.369    7.97
   43.42   7.784  44.665   7.617  46.342    8.32  47.684   8.725  47.865   9.211
  49.631   10.12  53.068  10.293      58  12.763   62.74  12.938
#Mann= 3 , 0 , 0
       0    .035       0       0    .035       0   62.74    .035       0
Bank Sta=0,62.74
XS Rating Curve= 0
Exp/Cntr=.3,.1

Type RM Length L Ch R = 1 ,395.5   ,7.34,7.34,7.34
XS GIS Cut Line= 2
      1616055.12      4854905.96 1616072.0293567 4854952.9482125
#Sta/Elev= 23
       0  12.757   3.784  12.717   6.564  13.525   7.962  13.659   9.085  13.582
   12.04  11.589  17.552  10.895  20.691   9.372   21.14   8.894  22.385    8.47
  23.972   8.514  26.467   8.298  28.917   8.322  30.762   8.374  34.001   8.313
  35.965   8.546  36.628   8.769  37.537   9.795   39.29   10.27  43.183  10.572
  46.712  13.424  47.219   13.74  50.028  13.702
#Mann= 3 , 0 , 0
       0    .035       0       0    .035       0  50.028    .035       0
Bank Sta=0,50.028
XS Rating Curve= 0
Exp/Cntr=.3,.1

Type RM Length L Ch R = 1 ,395     ,16.01,16.01,16.01
XS GIS Cut Line= 3
      1616047.58      4854906.69      1616065.94      4854955.36
 1616065.9410946 4854955.3629018
#Sta/Elev= 19
       0  14.195  10.841  14.093  11.801  13.854  16.634  10.521  21.487  10.161
  22.447   9.028    23.8   8.699  24.652   8.954  25.944    8.74  28.788   8.661
   31.11   8.393  33.988   8.611  35.249   8.524  37.958   8.508  39.975   8.775
  41.282  10.223  43.303  10.408  49.004  14.029  52.283    14.1
#Mann= 3 , 0 , 0
       0    .035       0       0    .035       0  52.283    .035       0
Bank Sta=0,52.283
XS Rating Curve= 0
Exp/Cntr=.3,.1

Type RM Length L Ch R = 1 ,394     ,6,6,6
XS GIS Cut Line= 3
      1616042.47      4854904.37      1616066.52      4854969.77
 1616067.1464286 4854971.4734691
#Sta/Elev= 27
       0  14.212   6.101  14.279   11.92  13.214  12.044  10.577  13.993  10.344
  16.677   10.07   18.09   8.789  19.886   8.816  20.439   8.845  21.799   8.595
  22.304    8.61  23.287    8.65  24.885   8.473  26.366   8.591   28.54   8.594
  30.113    8.77  30.734   8.752  32.147     8.8  32.828   8.851  34.419   8.749
  36.188   8.618  36.934   8.918  38.789    10.2  40.655  10.477  40.655  13.264
  46.566  14.284  53.745  14.319
#Mann= 3 , 0 , 0
       0    .035       0       0    .035       0  53.745    .035       0
Bank Sta=0,53.745
XS Rating Curve= 0
Exp/Cntr=.3,.1

Type RM Length L Ch R = 3 ,393.7   ,,,
BEGIN DESCRIPTION:
Ponte di Montuolo
END DESCRIPTION:
Bridge Culvert--1,0,-1,-1, 0
Deck Dist Width WeirC Skew NumUp NumDn MinLoCord MaxHiCord MaxSubmerge Is_Ogee
.5,5,1.44,0, 20, 20, , , .95, 0, 0,0,,
     6.1   11.92   19.89   19.89   20.44   20.44    21.8    21.8    22.3    22.3
   30.11   30.11   30.73   30.73   32.15   32.15   32.83   32.83   40.66   46.57
   14.28   14.28   14.28   14.28   14.28   14.28   14.28   14.28   14.28   14.28
   14.28   14.28   14.28   14.28   14.28   14.28   14.28   14.28   14.28   14.28
   14.28   13.21   13.21    8.81    8.84   13.21   13.21     8.6    8.61   13.21
   13.21    8.77    8.75   13.21   13.21     8.8    8.85   13.21   13.21   14.28
     6.1   11.92   19.89   19.89   20.44   20.44    21.8    21.8    22.3    22.3
   30.11   30.11   30.73   30.73   32.15   32.15   32.83   32.83   40.66   46.57
   14.28   14.28   14.28   14.28   14.28   14.28   14.28   14.28   14.28   14.28
   14.28   14.28   14.28   14.28   14.28   14.28   14.28   14.28   14.28   14.28
   14.28   13.21   13.21    8.81    8.84   13.21   13.21     8.6    8.61   13.21
   13.21    8.77    8.75   13.21   13.21     8.8    8.85   13.21   13.21   14.28
BR Coef=-1 , 0 , 0 ,1.25, 0 ,,,.8,-1,2,0,
WSPro=,,,, 1 ,,,, 0 ,,,, 0 ,,,,-1 ,-1 ,-1 , 0 , 0 , 0 , 0 , 0
BC Design=,, 0 ,, 0 ,,,,,,
BC HTab Sub Flow Pts= 40

Type RM Length L Ch R = 1 ,393     ,1,1,1
XS GIS Cut Line= 3
      1616040.42      4854911.21      1616061.21      4854967.87
 1616061.8369332 4854969.5786116
#Sta/Elev= 27
       0   14.21     6.1   14.28   11.92   13.21   12.04   10.58   13.99   10.34
   16.68   10.07   18.09    8.79   19.89    8.81   20.44    8.84    21.8     8.6
    22.3    8.61   23.29    8.65   24.89    8.47   26.37    8.59   28.54    8.59
   30.11    8.77   30.73    8.75   32.15     8.8   32.83    8.85   34.42    8.75
   36.19    8.62   36.93    8.92   38.79    10.2   40.66   10.48    40.8   13.26
   46.57   14.28   53.75   14.32
#Mann= 3 , 0 , 0
       0    .035       0       0    .035       0   53.75    .035       0
Bank Sta=0,53.75
XS Rating Curve= 0
Exp/Cntr=.3,.1

Type RM Length L Ch R = 1 ,392     ,46.38,46.38,46.38
XS GIS Cut Line= 3
      1616036.33       4854916.3 1616047.2194381 4854958.0943823
 1616047.2204461  4854958.098251
#Sta/Elev= 19
       0  14.163   5.174  13.844   9.567  10.935   13.35  10.505  16.352   10.07
   17.77   8.978  18.757   8.737  21.263   8.583  24.061   8.368  25.599   8.343
  27.013   8.426  28.915   8.401  32.501   8.668  33.524   9.209  35.112  10.055
  40.044  10.487  44.189  13.714  48.231  13.776  51.934  13.625
#Mann= 3 , 0 , 0
       0    .035       0       0    .035       0  51.934    .035       0
Bank Sta=0,51.934
XS Rating Curve= 0
Exp/Cntr=.3,.1

Type RM Length L Ch R = 1 ,391     ,46.59,46.59,46.59
XS GIS Cut Line= 2
       1616003.3      514854920.7541616005.998184814854970.99896
#Sta/Elev= 16
       0  13.766   4.404   13.33   8.222  11.175  11.566  10.819  14.692  10.598
  16.927   9.955  18.549   9.294  20.968   8.603  23.159   7.924  26.569   7.993
  29.615   8.074  32.698   8.531  33.801   9.575  38.983  10.203  44.575  13.079
  51.588  13.199
#Mann= 3 , 0 , 0
       0    .035       0       0    .035       0  51.588    .035       0
Bank Sta=0,51.588
XS Rating Curve= 0
Exp/Cntr=.3,.1

Type RM Length L Ch R = 1 ,390     ,13.47,13.47,13.47
XS GIS Cut Line= 2
      1615971.55      4854906.07 1615973.0885039 4854902.3636043
#Sta/Elev= 17
       0  13.699   5.318  13.458   9.804  11.425  13.697  11.089  17.686  10.647
  22.475   9.183  26.058   8.805  28.435   8.011  31.204   7.021  33.372   6.851
  35.548   8.101  37.856   8.607  39.569  10.005   43.43  10.137  49.188  13.086
  52.654   12.72  60.996   12.72
#Mann= 3 , 0 , 0
       0    .035       0       0    .035       0  60.996    .035       0
Bank Sta=0,60.996
XS Rating Curve= 0
Exp/Cntr=.3,.1

Type RM Length L Ch R = 1 ,389     ,10.63,10.63,10.63
XS GIS Cut Line= 2
      1615963.77      4854897.38      1615926.72      4854974.21
#Sta/Elev= 18
       0  13.587   4.482   13.57   9.869  13.264  13.164  11.704  16.724  11.105
  20.579  10.751   25.14   9.489  27.816   9.155  30.916     8.6  33.097   8.056
  35.819   6.987  39.087    6.46  42.084    7.28  45.218   8.292  49.427   8.556
  59.294   8.888  65.077   8.854   85.38   8.931
#Mann= 3 , 0 , 0
       0    .035       0       0    .035       0   85.38    .035       0
Bank Sta=0,85.38
XS Rating Curve= 0
Exp/Cntr=.3,.1

Type RM Length L Ch R = 1 ,388     ,22.24,22.24,22.24
XS GIS Cut Line= 2
      1615960.46      4854895.78 1615946.5352488 4854914.6378724
#Sta/Elev= 19
       0   13.65   5.662  13.548   9.824  13.191  13.384  11.249  17.777  10.941
  19.983  10.688  23.862   9.694   25.26   9.191  28.585   8.572  31.405   8.211
  34.073   7.611  36.489   7.801  39.268   7.751  41.926   8.514  43.411   9.868
  46.495  10.205   48.25  10.559  52.449  12.612  61.222  12.479
#Mann= 3 , 0 , 0
       0    .035       0       0    .035       0  61.222    .035       0
Bank Sta=0,61.222
XS Rating Curve= 0
Exp/Cntr=.3,.1

Type RM Length L Ch R = 1 ,387     ,65.15,65.15,65.15
XS GIS Cut Line= 2
      1615944.29      4854875.38 1615904.3505468 4854936.4891634
#Sta/Elev= 20
       0  13.588  11.151  13.483  18.179  13.359  22.657  11.324  26.323  10.913
   29.86  10.027  31.097   9.341  34.027    8.62   36.43   8.375  38.817   8.321
  41.988   7.528  45.007   7.841  48.904   8.361  49.607   9.315  54.598  10.055
  57.242  10.425  60.953   12.42  62.954  12.521  64.339  12.149  73.059  12.149
#Mann= 3 , 0 , 0
       0    .035       0       0    .035       0  73.059    .035       0
Bank Sta=0,73.059
XS Rating Curve= 0
Exp/Cntr=.3,.1

Type RM Length L Ch R = 1 ,386     ,57.45,57.45,57.45
XS GIS Cut Line= 2
      1615879.77      4854846.42      1615853.62      4854902.06
#Sta/Elev= 16
       0  13.164  14.872  12.998  19.251  10.585   22.08   10.27  25.732   9.971
  27.088   8.561  30.278   7.815  32.936   7.742   35.76   7.989  39.281     8.1
  42.651   8.486  44.679   9.806  48.641  10.018  52.437  10.323  55.102   11.98
   61.49   12.13
#Mann= 3 , 0 , 0
       0    .035       0       0    .035       0   61.49    .035       0
Bank Sta=0,61.49
XS Rating Curve= 0
Exp/Cntr=.3,.1

Type RM Length L Ch R = 1 ,385     ,32.12,32.12,32.12
XS GIS Cut Line= 3
      1615819.24      4854831.16      1615801.41      4854889.98
 1615801.4097388 4854889.9808616
#Sta/Elev= 24
       0  13.303   2.039  12.919   3.466  13.144   8.009  12.909   9.108   12.77
  13.211  10.327  19.414   9.912  20.771    8.33  24.693   7.397   26.41   7.475
  28.445   7.775  30.502   7.985  32.148   8.194  35.144   8.461  37.083   9.386
  38.385   9.714  47.885  10.566  50.609  11.207  50.694  12.877  52.641  12.792
  52.853  11.352  54.073   11.55  55.472  11.969  61.611  11.982
#Mann= 3 , 0 , 0
       0    .035       0       0    .035       0  61.611    .035       0
Bank Sta=0,61.611
XS Rating Curve= 0
Exp/Cntr=.3,.1

Type RM Length L Ch R = 1 ,384     ,49.95,49.95,49.95
XS GIS Cut Line= 2
      1615789.14      4854821.39 1615771.4127451  4854877.431322
#Sta/Elev= 21
       0  13.394.8329999  13.242   1.446  12.993   2.087  12.955    3.04   13.13
   7.813  12.863  13.408  10.194  20.413   9.799  21.383   8.435   25.01   7.566
  26.811   7.408   29.49    7.44  31.496   7.811  33.476   8.126  34.878   8.324
  35.162   8.825  39.432   9.627  45.554  10.254  49.393   12.29  51.464  12.313
  58.931  12.076
#Mann= 3 , 0 , 0
       0    .035       0       0    .035       0  58.931    .035       0
Bank Sta=0,58.931
XS Rating Curve= 0
Exp/Cntr=.3,.1

Type RM Length L Ch R = 1 ,383     ,48.12,48.12,48.12
XS GIS Cut Line= 2
      1615741.66      4854806.35   1615722.23096 4854863.9171555
#Sta/Elev= 19
       0  13.463    .666  13.358   1.223  13.043   1.785  13.061   2.221  13.214
   6.089  13.119  11.764  10.262  19.152   9.752  20.474    8.46  23.927   7.792
  26.122   7.492  29.191    7.56  32.102   7.911  35.544   8.295  37.387   8.503
  40.323    9.92  45.856  10.384  49.983  12.527  60.807  12.685
#Mann= 3 , 0 , 0
       0    .035       0       0    .035       0  60.807    .035       0
Bank Sta=0,60.807
XS Rating Curve= 0
Exp/Cntr=.3,.1

Type RM Length L Ch R = 1 ,382     ,56.96,56.96,56.96
XS GIS Cut Line= 2
      1615697.89      4854790.78 1615678.8018268 4854839.4253445
#Sta/Elev= 18
       0  13.805    .842  13.643   2.658  13.618   4.058  13.699   6.805  13.662
  13.741  10.078  18.862   9.826  20.571   8.482  23.724   7.828   25.71   7.658
  27.942   7.411   29.97   7.497  31.947   8.455  35.216   8.545  39.002   9.967
  45.629  10.717  49.924  13.138  52.285  13.162
#Mann= 3 , 0 , 0
       0    .035       0       0    .035       0  52.285    .035       0
Bank Sta=0,52.285
XS Rating Curve= 0
Exp/Cntr=.3,.1

Type RM Length L Ch R = 1 ,381     ,42.92,42.92,42.92
XS GIS Cut Line= 2
      1615655.02      4854742.67 1615624.8100354 4854821.6399074
#Sta/Elev= 27
       0  13.709   1.587  13.174   2.783  13.234  13.804  13.237  21.478  13.218
  27.165  13.155  29.452   12.99  32.636  12.611  35.627  12.518  39.609  12.589
  44.402  10.047  49.177    9.88  51.457   8.542  53.261   8.257  55.133   7.399
  57.161   7.368  59.206    7.17  61.106   7.533  62.677       8  64.788   8.475
  65.534   8.943  70.474   9.977   81.22  11.031  81.326   12.94   83.35  12.929
   83.43  10.983   84.72  11.429
#Mann= 3 , 0 , 0
       0    .035       0       0    .035       0   84.72    .035       0
Bank Sta=0,84.72
XS Rating Curve= 0
Exp/Cntr=.3,.1

Type RM Length L Ch R = 1 ,380     ,49.04,49.04,49.04
XS GIS Cut Line= 2
      1615609.32      4854740.86 1615583.6502837 4854808.6592508
#Sta/Elev= 20
       0  12.025   6.702  11.937  16.603  11.962  21.596  11.996  23.362  12.324
  31.184   9.976  35.809   9.689  37.422   8.345  39.484   8.001  42.495   7.961
  45.424   7.654  48.447   7.688  50.528    8.35   52.74   8.431   54.99   9.673
  64.002  10.414  68.532  12.854  69.608  12.848  70.431  12.564  72.519  12.458
#Mann= 3 , 0 , 0
       0    .035       0       0    .035       0  72.519    .035       0
Bank Sta=0,72.519
XS Rating Curve= 0
Exp/Cntr=.3,.1

Type RM Length L Ch R = 1 ,379     ,56.91,56.91,56.91
XS GIS Cut Line= 3
      1615559.37      4854729.63      1615536.39      4854800.39
 1615536.3884565 4854800.3947529
#Sta/Elev= 20
       0  12.653   4.455  12.476   9.112  12.665  13.905  12.406  17.974  12.496
   21.14  12.421  25.279  10.205  29.344   9.982  30.998   8.398  32.877   8.031
  35.052   7.853  37.106    7.73  40.138   7.603  44.103    8.32  46.732   8.696
  48.855    9.74  58.157  10.432  63.272  12.839  66.066  12.671  74.435  12.449
#Mann= 3 , 0 , 0
       0    .035       0       0    .035       0  74.435    .035       0
Bank Sta=0,74.435
XS Rating Curve= 0
Exp/Cntr=.3,.1

Type RM Length L Ch R = 1 ,378     ,46.06,46.06,46.06
XS GIS Cut Line= 2
      1615506.83      4854713.79      1615479.65      4854785.38
#Sta/Elev= 22
       0  12.341   7.642  12.376   13.83  12.431  18.273   12.45  20.049   11.92
  20.126  11.185  22.788  10.552  27.664   9.967  28.099   9.356  29.685   9.038
  30.093   8.422  33.503   7.746  36.047    7.49  39.415   7.763   42.41   8.033
  44.381   8.607  44.891    9.12   46.29   9.382  55.717  10.339  60.161  12.862
  63.479  12.617   76.67  12.504
#Mann= 3 , 0 , 0
       0    .035       0       0    .035       0   76.67    .035       0
Bank Sta=0,76.67
XS Rating Curve= 0
Exp/Cntr=.3,.1

Type RM Length L Ch R = 1 ,377     ,46.66,46.66,46.66
XS GIS Cut Line= 2
      1615470.24      4854689.14 1615459.2208456 4854713.4166805
#Sta/Elev= 27
       0  12.318   9.459  12.412  17.069  12.496   23.45  12.682   26.66  12.537
   27.59  12.431  32.043  10.673  37.246  10.278  39.514   9.281  40.429   8.482
  42.425    8.36   44.59   7.905  47.546   7.435  49.597    7.51  53.331   8.101
  54.824   8.185  54.918    8.63  57.133   9.302  58.714   9.652  62.622   9.847
  64.786  10.102  68.787  12.503  71.234  12.928  72.201  13.278  73.956  13.022
  75.322  12.351  78.761  12.221
#Mann= 3 , 0 , 0
       0    .035       0       0    .035       0  78.761    .035       0
Bank Sta=0,78.761
XS Rating Curve= 0
Exp/Cntr=.3,.1

Type RM Length L Ch R = 1 ,376     ,54.28,54.28,54.28
XS GIS Cut Line= 2
      1615428.55      4854671.63    1615417.1289 4854694.7923895
#Sta/Elev= 25
       0  12.175  15.427   12.19  22.777  12.206  24.263   12.38  25.801  12.862
  26.315  12.267  29.253  10.798  35.983  10.293  40.375   8.981  40.811    8.46
   43.54   7.845  45.552   7.612  47.025   7.472  49.089   7.444   51.01   7.548
  53.272   8.146  55.012   8.245  56.811   9.169  57.574   9.598  61.914   9.943
  63.755  10.124  68.351  12.774  71.875  12.883  74.472  12.378   85.53  12.373
#Mann= 3 , 0 , 0
       0    .035       0       0    .035       0   85.53    .035       0
Bank Sta=0,85.53
XS Rating Curve= 0
Exp/Cntr=.3,.1

Type RM Length L Ch R = 1 ,375     ,49.86,49.86,49.86
XS GIS Cut Line= 2
      1615381.73      4854647.97 1615341.8347606 4854722.6310908
#Sta/Elev= 26
       0   9.888   9.135    9.92  18.748   9.897   23.12   9.855  25.223   9.777
  28.761   9.769  30.341    8.91  32.717   8.656   37.63    8.45  39.841   8.376
   41.62    8.31  42.931   8.094  44.635   7.926  46.764   7.943  49.688   7.506
  52.143   7.448  53.726   7.638  55.525   8.353  55.647   8.725  56.576   9.428
  58.279   9.987  62.629  10.364    64.3   10.61  68.099  12.879  71.719  12.719
   84.76  12.424
#Mann= 3 , 0 , 0
       0    .035       0       0    .035       0   84.76    .035       0
Bank Sta=0,84.76
XS Rating Curve= 0
Exp/Cntr=.3,.1

Type RM Length L Ch R = 1 ,374     ,44.24,44.24,44.24
XS GIS Cut Line= 2
      1615340.22      4854625.92 1615328.2537082 4854645.2376911
#Sta/Elev= 27
       0  12.183  16.272  12.389  19.707  12.251  21.545   12.69  22.735  12.767
  24.967  12.338  28.542  10.518   33.27  10.312  36.836   8.902  37.835   8.379
  39.089   8.305  45.086   7.581  47.084    7.49  52.123   7.984  53.528   8.323
  53.602   8.717  54.395   8.916  55.446   9.684  56.581   9.941  60.282  10.077
  62.429  10.255  67.034  12.965  68.038   12.85  69.776  12.207  78.095  12.117
  80.689  12.732   91.15  12.809
#Mann= 3 , 0 , 0
       0    .035       0       0    .035       0   91.15    .035       0
Bank Sta=0,91.15
XS Rating Curve= 0
Exp/Cntr=.3,.1

Type RM Length L Ch R = 1 ,373     ,55.42,55.42,55.42
XS GIS Cut Line= 2
      1615303.62      4854597.19 1615301.7812554  4854600.448899
#Sta/Elev= 17
       0  13.699   5.318  13.458   9.804  11.425  13.697  11.089  17.686  10.647
  22.475   9.183  26.058   8.805  28.435   8.011  31.204   7.021  33.372   6.851
  35.548   8.101  37.856   8.607  39.569  10.005   43.43  10.137  49.188  13.086
  52.654   12.72  60.996   12.72
#Mann= 3 , 0 , 0
       0    .035       0       0    .035       0  60.996    .035       0
Bank Sta=0,60.996
XS Rating Curve= 0
Exp/Cntr=.3,.1

Type RM Length L Ch R = 1 ,372     ,51.99,51.99,51.99
XS GIS Cut Line= 2
      1615257.42      4854572.62 1615241.7185745 4854597.1638073
#Sta/Elev= 29
       0  12.432   8.482  12.379  17.164  12.423  24.198   12.05  26.087  12.779
  29.137  12.929  30.527  12.772  34.475  10.107  38.782   9.801  41.815   8.882
  44.074    8.58  46.018   8.388  47.314   8.217  48.718   7.985    50.4   7.372
  51.952   6.928  53.023   6.888  54.184   6.864  55.476   7.154  57.554   7.886
  58.822   8.343  60.561   9.906   61.19  10.049  64.718  10.407  66.869  10.682
   70.85    12.9  72.978  12.891  75.025  12.223   77.61  12.059
#Mann= 3 , 0 , 0
       0    .035       0       0    .035       0   77.61    .035       0
Bank Sta=0,77.61
XS Rating Curve= 0
Exp/Cntr=.3,.1
